--- Corner_Brook2.prj (project) ---

Proj Title=Corner_Brook2
Current Plan=p18
Default Exp/Contr=0.3,0.1
SI Units
Geom File=g01
Geom File=g02
Geom File=g03
Flow File=f01
Flow File=f02
Flow File=f03
Flow File=f04
Plan File=p18
Plan File=p19
Y Axis Title=Elevation
X Axis Title(PF)=Main Channel Distance
X Axis Title(XS)=Station
BEGIN DESCRIPTION:
END DESCRIPTION:
DSS File=dss
DSS Export Rating Curves= 0
DSS Export Rating Curve Sorted= 0
DSS Export Volume Flow Curves= 0
DXF OffsetX= 0
DXF OffsetY= 0
DXF ScaleX= 1
DXF ScaleY= 10

--- Corner_Brook2.p18 (plan) ---

Plan Title=Plan 18
Program Version=5.01
Short Identifier=Plan 18
Geom File=g01
Flow File=f01
Mixed Flow
K Sum by GR= 0
Std Step Tol= 0.01
Critical Tol= 0.01
Num of Std Step Trials= 20
Max Error Tol= 0.3
Flow Tol Ratio= 0.001
Split Flow NTrial= 30
Split Flow Tol= 0.02
Split Flow Ratio= 0.02
Log Output Level= 0
Friction Slope Method= 1
Unsteady Friction Slope Method= 2
Unsteady Bridges Friction Slope Method= 1
Parabolic Critical Depth
Global Vel Dist= 0 , 0 , 0
Global Log Level= 0
CheckData=True
Encroach Param=-1 ,0,0, 0
Computation Interval=1HOUR
Output Interval=1HOUR
Instantaneous Interval=1HOUR
Mapping Interval=1HOUR
Run HTab= 0
Run UNet= 0
Run Sediment= 0
Run PostProcess= 0
Run WQNet= 0
Run RASMapper= 0
UNET Theta= 1
UNET Theta Warmup= 1
UNET ZTol= 0.02
UNET ZSATol= 0.05
UNET MxIter= 20
UNET Max Iter WO Improvement= 0
UNET MaxInSteps= 0
UNET DtIC= 0
UNET DtMin= 0
UNET MaxCRTS= 20
UNET WFStab= 2
UNET SFStab= 1
UNET WFX= 1
UNET SFX= 1
UNET DSS MLevel= 4
UNET Pardiso=0
UNET DZMax Abort= 100
UNET Use Existing IB Tables=-1
UNET Froude Reduction=False
UNET Froude Limit= 1
UNET Froude Power= 10
UNET Time Slicing=0,0, 5
UNET Junction Losses=0
UNET D1 Cores= 0
UNET D2 Coriolis=0
UNET D2 Cores= 0
UNET D2 Theta= 1
UNET D2 Theta Warmup= 1
UNET D2 Z Tol= 0.003
UNET D2 Volume Tol= 0.003
UNET D2 Max Iterations= 20
UNET D2 Equation= 0
UNET D2 RampUpFraction=0.1
UNET D2 TimeSlices= 1
UNET D2 BCVolumeCheck=0
UNET D1D2 MaxIter= 0
UNET D1D2 ZTol=0.003
UNET D1D2 QTol=0.1
UNET D1D2 MinQTol=0.03
DSS File=dss
Write IC File= 0
Write IC File at Fixed DateTime=0
Write IC File at Sim End=0
Echo Input=False
Echo Parameters=False
Echo Output=False
Write Detailed= 0
HDF Write Warmup=0
HDF Write Time Slices=0
HDF Flush=0
HDF Face Node Velocities=0
HDF Compression= 1
HDF Chunk Size= 1
HDF Spatial Parts= 1
HDF Use Max Rows=0
HDF Fixed Rows= 1
Calibration Method= 0
Calibration Iterations= 20
Calibration Max Change=0.05
Calibration Tolerance=0.2
Calibration Maximum=1.5
Calibration Minimum=0.5
Calibration Optimization Method= 1
WQ AD Non Conservative
WQ ULTIMATE=-1
WQ Max Comp Step=1HOUR
WQ Output Interval=15MIN
WQ Output Selected Increments= 0
WQ Output face flow=0
WQ Output face velocity=0
WQ Output face area=0
WQ Output face dispersion=0
WQ Output cell volume=0
WQ Output cell surface area=0
WQ Output cell continuity=0
WQ Output cumulative cell continuity=0
WQ Output face conc=0
WQ Output face dconc_dx=0
WQ Output face courant=0
WQ Output face peclet=0
WQ Output face adv mass=0
WQ Output face disp mass=0
WQ Output cell mass=0
WQ Output cell source sink temp=0
WQ Output nsm pathways=0
WQ Output nsm derived pathways=0
WQ Output MaxMinRange=-1
WQ Daily Max Min Mean=-1
WQ Daily Range=0
WQ Daily Time=0
WQ Create Restart=0
WQ Fixed Restart=0
WQ System Summary=0
WQ Write To DSS=0
WQ Use Fixed Temperature=0
Sorting and Armoring Iterations= 10
XS Update Threshold= 0.02
Bed Roughness Predictor= 0
Hydraulics Update Threshold= 0.02
Energy Slope Method= 1
Volume Change Method= 0
Sediment Retention Method= 0
XS Weighting Method= 0
Number of US Weighted Cross Sections= 1
Number of DS Weighted Cross Sections= 1
Upstream XS Weight=0.25
Main XS Weight=0.5
Downstream XS Weight=0.25
Number of DS XS's Weighted with US Boundary= 1
Upstream Boundary Weight= 1
Weight of XSs Associated with US Boundary= 0
Number of US XS's Weighted with DS Boundary= 1
Downstream Boundary Weight= 0.5
Weight of XSs Associated with DS Boundary= 0.5
Percentile Method= 0
Sediment Output Level= 4
Mass or Volume Output= 0
Output Increment Type= 1
Profile and TS Output Increment= 10
XS Output Flag= 0
XS Output Increment= 10
Write Gradation File= 0
Read Gradation Hotstart= 0
Write HDF5 File= 1
Write DSS Sediment File= 0
SV Curve= 0
Specific Gage Flag= 0

--- Corner_Brook2.p19 (plan) ---

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Plan Title=Plan 19
Program Version=4.10
Geom File=g02
Flow File=f03
UNET Convert EG Bridges= 0
WQ Output cell source sink nsm=0
Disregard all LS=0
Disregard all Conn=0
Disregard all Breaches=0
Disregard all Pumps=0

--- Corner_Brook2.f01 (steady flow) ---

Flow Title=20yr
Program Version=4.10
Number of Profiles= 25
Profile Names=20Year-Existing,FINIIS-20yr-2050-90%,FINIIS-20yr-2050-Max,AMEC-20yr-2020-90%,AMEC-20yr-2020-Max,AMEC-20yr-2050-90%,AMEC-20yr-2050-Max,AMEC-20yr-2080-90%,AMEC-20yr-2080-Max,CGCM2-20yr-2020-90%,CGCM2-20yr-2020-Max,CGCM2-20yr-2050-90%,CGCM2-20yr-2050-Max,CGCM2-20yr-2080-90%,CGCM2-20yr-2080-Max,HADCM3-20yr-2020-90%,HADCM3-20yr-2020-Max,HADCM3-20yr-2050-90%,HADCM3-20yr-2050-Max,HADCM3-20yr-2080-90%,HADCM3-20yr-2080-Max,PF 22,PF 23,PF 24,PF 25
River Rch & RM=BellsB,TR001           ,178.13
    12.5    29.2    28.6    13.8    14.8    14.3      15    14.9      16    20.6
    19.7    21.3    20.9    25.3    25.4    16.8    16.1    26.6    26.1    19.3
    19.4    12.5    12.5    12.5    12.5
River Rch & RM=BellsB,M002            ,5166.11
    10.4    23.6    23.1    11.4    12.2    11.8    12.3    12.3    13.1    16.9
    16.1    17.4      17    20.5    20.6    13.8    13.2    21.6    21.1    15.8
    15.9    10.4    10.4    10.4    10.4
River Rch & RM=BellsB,M002            ,4436.28
    18.8    41.9      41    20.6    21.9    21.4    22.2    22.2    23.7    30.4
      29      31    30.6    36.3    36.4      25    23.8    38.3    37.4    28.5
    28.6    18.8    18.8    18.8    18.8
River Rch & RM=BellsB,M002            ,3329.08
    23.8    52.3    51.1    25.9    27.5    26.8      28    27.9    29.8    38.5
    36.7    39.7    38.9    45.1    45.2    31.5      30    47.6    46.5    36.1
    36.2    23.8    23.8    23.8    23.8
River Rch & RM=BellsB,M002            ,2295.83
      26      56    54.8    27.8    29.6    28.8    30.1      30    32.1    41.6
    39.6    42.9      42    48.4    48.5    33.9    32.3    50.9    49.8    38.9
      39      26      26      26      26
River Rch & RM=BellsB,M001            ,1582.05
    41.3    90.2    88.3    44.7    47.3      46      48    47.9    51.3    66.4
    63.3    68.5    67.1    78.9    79.3    54.1    51.6    82.7    81.2    62.1
    62.4    41.3    41.3    41.3    41.3
River Rch & RM=BellsB,M001            ,816.09
    42.5    92.2    90.4    46.1    48.4    47.4    49.2      49    52.6      68
    64.8    70.2    68.7    80.8    81.2    55.3    52.8    84.8    83.2    63.6
    63.9    42.5    42.5    42.5    42.5
River Rch & RM=CornerB,M004            ,2888.71
   134.2   317.3   313.2   149.6   162.2   155.6   163.7   160.8   172.6   223.5
   216.8   231.3   228.3   272.5   274.4   182.3   176.7   289.3   285.7   208.2
   209.6   134.2   134.2   134.2   134.2
River Rch & RM=CornerB,TR001           ,206.04
    22.9    53.3    52.4    25.4    27.3    26.4    27.6    27.4    29.4    37.8
    36.3      39    38.4    46.1    46.5    30.9    29.7    48.7    47.9    35.3
    35.6    22.9    22.9    22.9    22.9
River Rch & RM=CornerB,M003            ,2689.92
   146.5   350.4   345.9   163.5   177.5   170.2   179.3     176     189   245.6
   238.2   254.3   251.1   300.3   302.4   199.8   193.7   319.1   315.1   228.6
   230.2     100      75      50      25
River Rch & RM=CornerB,M003            ,2267.71
   146.8   351.1   346.6   163.8   177.9   170.5   179.7   176.3   189.4   246.1
   238.7   254.8   251.5   300.9     303   200.2   194.1   319.7   315.7   229.1
   230.7     100      75      50      25
River Rch & RM=CornerB,TR002           ,21.04
     8.7    19.5    19.1     9.6    10.1     9.9    10.3    10.3      11      14
    13.4    14.4    14.1      17      17    11.5      11    17.9    17.5    13.1
    13.2     8.7     8.7     8.7     8.7
River Rch & RM=CornerB,M002            ,1826.39
   148.2   354.7   350.2   165.5   179.8   172.2   181.5   178.1   191.3   248.6
   241.2   257.4   254.2   303.9   306.1   202.2   196.2     323     319   231.4
     233     100      75      50      25
River Rch & RM=CornerB,M002            ,1539.91
   147.1   353.8   349.4   164.3   178.6     171   180.3   176.8   190.1   247.6
   240.2   256.4   253.3   302.9     305   201.1   195.2   322.1   318.1   230.3
   231.9     100      75      50      25
River Rch & RM=CornerB,M002            ,915.75
   146.2   353.2   348.8   163.5   177.9   170.2   179.5   175.9   189.2   246.8
   239.5   255.7   252.5   302.1   304.2   200.3   194.4   321.5   317.5   229.4
     231     100      75      50      25
River Rch & RM=CornerB,M002            ,828.33
   141.5   346.3     342   158.5   172.7   165.1   174.3   170.6   183.7   240.7
   233.6   249.5   246.5   295.4   297.4   194.7     189   314.7   310.9   223.4
     225     100      75      50      25
River Rch & RM=CornerB,M001            ,659.37
   148.4   365.9   361.6   166.6   182.1   173.7   183.6   179.4   193.2   253.8
   246.8   263.3   260.2   311.7   313.8   205.1   199.4   332.4   328.5   235.4
     237     100      75      50      25
Boundary for River Rch & Prof#=BellsB,TR001           , 1
Up Type= 3
Up Slope=0.043
Dn Type= 0
Boundary for River Rch & Prof#=BellsB,TR001           , 2
Up Type= 3
Up Slope=0.043
Dn Type= 0
Boundary for River Rch & Prof#=BellsB,TR001           , 3
Up Type= 3
Up Slope=0.043
Dn Type= 0
Boundary for River Rch & Prof#=BellsB,TR001           , 4
Up Type= 3
Up Slope=0.043
Dn Type= 0
Boundary for River Rch & Prof#=BellsB,TR001           , 5
Up Type= 3
Up Slope=0.043
Dn Type= 0
Boundary for River Rch & Prof#=BellsB,TR001           , 6
Up Type= 3
Up Slope=0.043
Dn Type= 0
Boundary for River Rch & Prof#=BellsB,TR001           , 7
Up Type= 3
Up Slope=0.043
Dn Type= 0
Boundary for River Rch & Prof#=BellsB,TR001           , 8
Up Type= 3
Up Slope=0.043
Dn Type= 0
Boundary for River Rch & Prof#=BellsB,TR001           , 9
Up Type= 3
Up Slope=0.043
Dn Type= 0
Boundary for River Rch & Prof#=BellsB,TR001           , 10
Up Type= 3
Up Slope=0.043
Dn Type= 0
Boundary for River Rch & Prof#=BellsB,TR001           , 11
Up Type= 3
Up Slope=0.043
Dn Type= 0
Boundary for River Rch & Prof#=BellsB,TR001           , 12
Up Type= 3
Up Slope=0.043
Dn Type= 0
Boundary for River Rch & Prof#=BellsB,TR001           , 13
Up Type= 3
Up Slope=0.043
Dn Type= 0
Boundary for River Rch & Prof#=BellsB,TR001           , 14
Up Type= 3
Up Slope=0.043
Dn Type= 0
Boundary for River Rch & Prof#=BellsB,TR001           , 15
Up Type= 3
Up Slope=0.043
Dn Type= 0
Boundary for River Rch & Prof#=BellsB,TR001           , 16
Up Type= 3
Up Slope=0.043
Dn Type= 0
Boundary for River Rch & Prof#=BellsB,TR001           , 17
Up Type= 3
Up Slope=0.043
Dn Type= 0
Boundary for River Rch & Prof#=BellsB,TR001           , 18
Up Type= 3
Up Slope=0.043
Dn Type= 0
Boundary for River Rch & Prof#=BellsB,TR001           , 19
Up Type= 3
Up Slope=0.043
Dn Type= 0
Boundary for River Rch & Prof#=BellsB,TR001           , 20
Up Type= 3
Up Slope=0.043
Dn Type= 0
Boundary for River Rch & Prof#=BellsB,TR001           , 21
Up Type= 3
Up Slope=0.043
Dn Type= 0
Boundary for River Rch & Prof#=BellsB,M002            , 1
Up Type= 3
Up Slope=0.013
Dn Type= 0
Boundary for River Rch & Prof#=BellsB,M002            , 2
Up Type= 3
Up Slope=0.013
Dn Type= 0
Boundary for River Rch & Prof#=BellsB,M002            , 3
Up Type= 3
Up Slope=0.013
Dn Type= 0
Boundary for River Rch & Prof#=BellsB,M002            , 4
Up Type= 3
Up Slope=0.013
Dn Type= 0
Boundary for River Rch & Prof#=BellsB,M002            , 5
Up Type= 3
Up Slope=0.013
Dn Type= 0
Boundary for River Rch & Prof#=BellsB,M002            , 6
Up Type= 3
Up Slope=0.013
Dn Type= 0
Boundary for River Rch & Prof#=BellsB,M002            , 7
Up Type= 3
Up Slope=0.013
Dn Type= 0
Boundary for River Rch & Prof#=BellsB,M002            , 8
Up Type= 3
Up Slope=0.013
Dn Type= 0
Boundary for River Rch & Prof#=BellsB,M002            , 9
Up Type= 3
Up Slope=0.013
Dn Type= 0
Boundary for River Rch & Prof#=BellsB,M002            , 10
Up Type= 3
Up Slope=0.013
Dn Type= 0
Boundary for River Rch & Prof#=BellsB,M002            , 11
Up Type= 3
Up Slope=0.013
Dn Type= 0
Boundary for River Rch & Prof#=BellsB,M002            , 12
Up Type= 3
Up Slope=0.013
Dn Type= 0
Boundary for River Rch & Prof#=BellsB,M002            , 13
Up Type= 3
Up Slope=0.013
Dn Type= 0
Boundary for River Rch & Prof#=BellsB,M002            , 14
Up Type= 3
Up Slope=0.013
Dn Type= 0
Boundary for River Rch & Prof#=BellsB,M002            , 15
Up Type= 3
Up Slope=0.013
Dn Type= 0
Boundary for River Rch & Prof#=BellsB,M002            , 16
Up Type= 3
Up Slope=0.013
Dn Type= 0
Boundary for River Rch & Prof#=BellsB,M002            , 17
Up Type= 3
Up Slope=0.013
Dn Type= 0
Boundary for River Rch & Prof#=BellsB,M002            , 18
Up Type= 3
Up Slope=0.013
Dn Type= 0
Boundary for River Rch & Prof#=BellsB,M002            , 19
Up Type= 3
Up Slope=0.013
Dn Type= 0
Boundary for River Rch & Prof#=BellsB,M002            , 20
Up Type= 3
Up Slope=0.013
Dn Type= 0
Boundary for River Rch & Prof#=BellsB,M002            , 21
Up Type= 3
Up Slope=0.013
Dn Type= 0
Boundary for River Rch & Prof#=BellsB,M001            , 1
Up Type= 0
Dn Type= 0
Boundary for River Rch & Prof#=BellsB,M001            , 2
Up Type= 0
Dn Type= 0
Boundary for River Rch & Prof#=BellsB,M001            , 3
Up Type= 0
Dn Type= 0
Boundary for River Rch & Prof#=BellsB,M001            , 4
Up Type= 0
Dn Type= 0
Boundary for River Rch & Prof#=BellsB,M001            , 5
Up Type= 0
Dn Type= 0
Boundary for River Rch & Prof#=BellsB,M001            , 6
Up Type= 0
Dn Type= 0
Boundary for River Rch & Prof#=BellsB,M001            , 7
Up Type= 0
Dn Type= 0
Boundary for River Rch & Prof#=BellsB,M001            , 8
Up Type= 0
Dn Type= 0
Boundary for River Rch & Prof#=BellsB,M001            , 9
Up Type= 0
Dn Type= 0
Boundary for River Rch & Prof#=BellsB,M001            , 10
Up Type= 0
Dn Type= 0
Boundary for River Rch & Prof#=BellsB,M001            , 11
Up Type= 0
Dn Type= 0
Boundary for River Rch & Prof#=BellsB,M001            , 12
Up Type= 0
Dn Type= 0
Boundary for River Rch & Prof#=BellsB,M001            , 13
Up Type= 0
Dn Type= 0
Boundary for River Rch & Prof#=BellsB,M001            , 14
Up Type= 0
Dn Type= 0
Boundary for River Rch & Prof#=BellsB,M001            , 15
Up Type= 0
Dn Type= 0
Boundary for River Rch & Prof#=BellsB,M001            , 16
Up Type= 0
Dn Type= 0
Boundary for River Rch & Prof#=BellsB,M001            , 17
Up Type= 0
Dn Type= 0
Boundary for River Rch & Prof#=BellsB,M001            , 18
Up Type= 0
Dn Type= 0
Boundary for River Rch & Prof#=BellsB,M001            , 19
Up Type= 0
Dn Type= 0
Boundary for River Rch & Prof#=BellsB,M001            , 20
Up Type= 0
Dn Type= 0
Boundary for River Rch & Prof#=BellsB,M001            , 21
Up Type= 0
Dn Type= 0
Boundary for River Rch & Prof#=CornerB,M004            , 1
Up Type= 3
Up Slope=0.006
Dn Type= 0
Boundary for River Rch & Prof#=CornerB,M004            , 2
Up Type= 3
Up Slope=0.006
Dn Type= 0
Boundary for River Rch & Prof#=CornerB,M004            , 3
Up Type= 3
Up Slope=0.006
Dn Type= 0
Boundary for River Rch & Prof#=CornerB,M004            , 4
Up Type= 3
Up Slope=0.006
Dn Type= 0
Boundary for River Rch & Prof#=CornerB,M004            , 5
Up Type= 3
Up Slope=0.006
Dn Type= 0
Boundary for River Rch & Prof#=CornerB,M004            , 6
Up Type= 3
Up Slope=0.006
Dn Type= 0
Boundary for River Rch & Prof#=CornerB,M004            , 7
Up Type= 3
Up Slope=0.006
Dn Type= 0
Boundary for River Rch & Prof#=CornerB,M004            , 8
Up Type= 3
Up Slope=0.006
Dn Type= 0
Boundary for River Rch & Prof#=CornerB,M004            , 9
Up Type= 3
Up Slope=0.006
Dn Type= 0
Boundary for River Rch & Prof#=CornerB,M004            , 10
Up Type= 3
Up Slope=0.006
Dn Type= 0
Boundary for River Rch & Prof#=CornerB,M004            , 11
Up Type= 3
Up Slope=0.006
Dn Type= 0
Boundary for River Rch & Prof#=CornerB,M004            , 12
Up Type= 3
Up Slope=0.006
Dn Type= 0
Boundary for River Rch & Prof#=CornerB,M004            , 13
Up Type= 3
Up Slope=0.006
Dn Type= 0
Boundary for River Rch & Prof#=CornerB,M004            , 14
Up Type= 3
Up Slope=0.006
Dn Type= 0
Boundary for River Rch & Prof#=CornerB,M004            , 15
Up Type= 3
Up Slope=0.006
Dn Type= 0
Boundary for River Rch & Prof#=CornerB,M004            , 16
Up Type= 3
Up Slope=0.006
Dn Type= 0
Boundary for River Rch & Prof#=CornerB,M004            , 17
Up Type= 3
Up Slope=0.006
Dn Type= 0
Boundary for River Rch & Prof#=CornerB,M004            , 18
Up Type= 3
Up Slope=0.006
Dn Type= 0
Boundary for River Rch & Prof#=CornerB,M004            , 19
Up Type= 3
Up Slope=0.006
Dn Type= 0
Boundary for River Rch & Prof#=CornerB,M004            , 20
Up Type= 3
Up Slope=0.006
Dn Type= 0
Boundary for River Rch & Prof#=CornerB,M004            , 21
Up Type= 3
Up Slope=0.006
Dn Type= 0
Boundary for River Rch & Prof#=CornerB,TR001           , 1
Up Type= 3
Up Slope=0.042
Dn Type= 0
Boundary for River Rch & Prof#=CornerB,TR001           , 2
Up Type= 3
Up Slope=0.042
Dn Type= 0
Boundary for River Rch & Prof#=CornerB,TR001           , 3
Up Type= 3
Up Slope=0.042
Dn Type= 0
Boundary for River Rch & Prof#=CornerB,TR001           , 4
Up Type= 3
Up Slope=0.042
Dn Type= 0
Boundary for River Rch & Prof#=CornerB,TR001           , 5
Up Type= 3
Up Slope=0.042
Dn Type= 0
Boundary for River Rch & Prof#=CornerB,TR001           , 6
Up Type= 3
Up Slope=0.042
Dn Type= 0
Boundary for River Rch & Prof#=CornerB,TR001           , 7
Up Type= 3
Up Slope=0.042
Dn Type= 0
Boundary for River Rch & Prof#=CornerB,TR001           , 8
Up Type= 3
Up Slope=0.042
Dn Type= 0
Boundary for River Rch & Prof#=CornerB,TR001           , 9
Up Type= 3
Up Slope=0.042
Dn Type= 0
Boundary for River Rch & Prof#=CornerB,TR001           , 10
Up Type= 3
Up Slope=0.042
Dn Type= 0
Boundary for River Rch & Prof#=CornerB,TR001           , 11
Up Type= 3
Up Slope=0.042
Dn Type= 0
Boundary for River Rch & Prof#=CornerB,TR001           , 12
Up Type= 3
Up Slope=0.042
Dn Type= 0
Boundary for River Rch & Prof#=CornerB,TR001           , 13
Up Type= 3
Up Slope=0.042
Dn Type= 0
Boundary for River Rch & Prof#=CornerB,TR001           , 14
Up Type= 3
Up Slope=0.042
Dn Type= 0
Boundary for River Rch & Prof#=CornerB,TR001           , 15
Up Type= 3
Up Slope=0.042
Dn Type= 0
Boundary for River Rch & Prof#=CornerB,TR001           , 16
Up Type= 3
Up Slope=0.042
Dn Type= 0
Boundary for River Rch & Prof#=CornerB,TR001           , 17
Up Type= 3
Up Slope=0.042
Dn Type= 0
Boundary for River Rch & Prof#=CornerB,TR001           , 18
Up Type= 3
Up Slope=0.042
Dn Type= 0
Boundary for River Rch & Prof#=CornerB,TR001           , 19
Up Type= 3
Up Slope=0.042
Dn Type= 0
Boundary for River Rch & Prof#=CornerB,TR001           , 20
Up Type= 3
Up Slope=0.042
Dn Type= 0
Boundary for River Rch & Prof#=CornerB,TR001           , 21
Up Type= 3
Up Slope=0.042
Dn Type= 0
Boundary for River Rch & Prof#=CornerB,M003            , 1
Up Type= 0
Dn Type= 0
Boundary for River Rch & Prof#=CornerB,M003            , 2
Up Type= 0
Dn Type= 0
Boundary for River Rch & Prof#=CornerB,M003            , 3
Up Type= 0
Dn Type= 0
Boundary for River Rch & Prof#=CornerB,M003            , 4
Up Type= 0
Dn Type= 0
Boundary for River Rch & Prof#=CornerB,M003            , 5
Up Type= 0
Dn Type= 0
Boundary for River Rch & Prof#=CornerB,M003            , 6
Up Type= 0
Dn Type= 0
Boundary for River Rch & Prof#=CornerB,M003            , 7
Up Type= 0
Dn Type= 0
Boundary for River Rch & Prof#=CornerB,M003            , 8
Up Type= 0
Dn Type= 0
Boundary for River Rch & Prof#=CornerB,M003            , 9
Up Type= 0
Dn Type= 0
Boundary for River Rch & Prof#=CornerB,M003            , 10
Up Type= 0
Dn Type= 0
Boundary for River Rch & Prof#=CornerB,M003            , 11
Up Type= 0
Dn Type= 0
Boundary for River Rch & Prof#=CornerB,M003            , 12
Up Type= 0
Dn Type= 0
Boundary for River Rch & Prof#=CornerB,M003            , 13
Up Type= 0
Dn Type= 0
Boundary for River Rch & Prof#=CornerB,M003            , 14
Up Type= 0
Dn Type= 0
Boundary for River Rch & Prof#=CornerB,M003            , 15
Up Type= 0
Dn Type= 0
Boundary for River Rch & Prof#=CornerB,M003            , 16
Up Type= 0
Dn Type= 0
Boundary for River Rch & Prof#=CornerB,M003            , 17
Up Type= 0
Dn Type= 0
Boundary for River Rch & Prof#=CornerB,M003            , 18
Up Type= 0
Dn Type= 0
Boundary for River Rch & Prof#=CornerB,M003            , 19
Up Type= 0
Dn Type= 0
Boundary for River Rch & Prof#=CornerB,M003            , 20
Up Type= 0
Dn Type= 0
Boundary for River Rch & Prof#=CornerB,M003            , 21
Up Type= 0
Dn Type= 0
Boundary for River Rch & Prof#=CornerB,TR002           , 1
Up Type= 3
Up Slope=0.15
Dn Type= 0
Boundary for River Rch & Prof#=CornerB,TR002           , 2
Up Type= 3
Up Slope=0.15
Dn Type= 0
Boundary for River Rch & Prof#=CornerB,TR002           , 3
Up Type= 3
Up Slope=0.15
Dn Type= 0
Boundary for River Rch & Prof#=CornerB,TR002           , 4
Up Type= 3
Up Slope=0.15
Dn Type= 0
Boundary for River Rch & Prof#=CornerB,TR002           , 5
Up Type= 3
Up Slope=0.15
Dn Type= 0
Boundary for River Rch & Prof#=CornerB,TR002           , 6
Up Type= 3
Up Slope=0.15
Dn Type= 0
Boundary for River Rch & Prof#=CornerB,TR002           , 7
Up Type= 3
Up Slope=0.15
Dn Type= 0
Boundary for River Rch & Prof#=CornerB,TR002           , 8
Up Type= 3
Up Slope=0.15
Dn Type= 0
Boundary for River Rch & Prof#=CornerB,TR002           , 9
Up Type= 3
Up Slope=0.15
Dn Type= 0
Boundary for River Rch & Prof#=CornerB,TR002           , 10
Up Type= 3
Up Slope=0.15
Dn Type= 0
Boundary for River Rch & Prof#=CornerB,TR002           , 11
Up Type= 3
Up Slope=0.15
Dn Type= 0
Boundary for River Rch & Prof#=CornerB,TR002           , 12
Up Type= 3
Up Slope=0.15
Dn Type= 0
Boundary for River Rch & Prof#=CornerB,TR002           , 13
Up Type= 3
Up Slope=0.15
Dn Type= 0
Boundary for River Rch & Prof#=CornerB,TR002           , 14
Up Type= 3
Up Slope=0.15
Dn Type= 0
Boundary for River Rch & Prof#=CornerB,TR002           , 15
Up Type= 3
Up Slope=0.15
Dn Type= 0
Boundary for River Rch & Prof#=CornerB,TR002           , 16
Up Type= 3
Up Slope=0.15
Dn Type= 0
Boundary for River Rch & Prof#=CornerB,TR002           , 17
Up Type= 3
Up Slope=0.15
Dn Type= 0
Boundary for River Rch & Prof#=CornerB,TR002           , 18
Up Type= 3
Up Slope=0.15
Dn Type= 0
Boundary for River Rch & Prof#=CornerB,TR002           , 19
Up Type= 3
Up Slope=0.15
Dn Type= 0
Boundary for River Rch & Prof#=CornerB,TR002           , 20
Up Type= 3
Up Slope=0.15
Dn Type= 0
Boundary for River Rch & Prof#=CornerB,TR002           , 21
Up Type= 3
Up Slope=0.15
Dn Type= 0
Boundary for River Rch & Prof#=CornerB,M002            , 1
Up Type= 0
Dn Type= 0
Boundary for River Rch & Prof#=CornerB,M002            , 2
Up Type= 0
Dn Type= 0
Boundary for River Rch & Prof#=CornerB,M002            , 3
Up Type= 0
Dn Type= 0
Boundary for River Rch & Prof#=CornerB,M002            , 4
Up Type= 0
Dn Type= 0
Boundary for River Rch & Prof#=CornerB,M002            , 5
Up Type= 0
Dn Type= 0
Boundary for River Rch & Prof#=CornerB,M002            , 6
Up Type= 0
Dn Type= 0
Boundary for River Rch & Prof#=CornerB,M002            , 7
Up Type= 0
Dn Type= 0
Boundary for River Rch & Prof#=CornerB,M002            , 8
Up Type= 0
Dn Type= 0
Boundary for River Rch & Prof#=CornerB,M002            , 9
Up Type= 0
Dn Type= 0
Boundary for River Rch & Prof#=CornerB,M002            , 10
Up Type= 0
Dn Type= 0
Boundary for River Rch & Prof#=CornerB,M002            , 11
Up Type= 0
Dn Type= 0
Boundary for River Rch & Prof#=CornerB,M002            , 12
Up Type= 0
Dn Type= 0
Boundary for River Rch & Prof#=CornerB,M002            , 13
Up Type= 0
Dn Type= 0
Boundary for River Rch & Prof#=CornerB,M002            , 14
Up Type= 0
Dn Type= 0
Boundary for River Rch & Prof#=CornerB,M002            , 15
Up Type= 0
Dn Type= 0
Boundary for River Rch & Prof#=CornerB,M002            , 16
Up Type= 0
Dn Type= 0
Boundary for River Rch & Prof#=CornerB,M002            , 17
Up Type= 0
Dn Type= 0
Boundary for River Rch & Prof#=CornerB,M002            , 18
Up Type= 0
Dn Type= 0
Boundary for River Rch & Prof#=CornerB,M002            , 19
Up Type= 0
Dn Type= 0
Boundary for River Rch & Prof#=CornerB,M002            , 20
Up Type= 0
Dn Type= 0
Boundary for River Rch & Prof#=CornerB,M002            , 21
Up Type= 0
Dn Type= 0
Boundary for River Rch & Prof#=CornerB,M001            , 1
Up Type= 0
Dn Type= 1
Dn Known WS=2.8
Boundary for River Rch & Prof#=CornerB,M001            , 2
Up Type= 0
Dn Type= 1
Dn Known WS=3.03
Boundary for River Rch & Prof#=CornerB,M001            , 3
Up Type= 0
Dn Type= 1
Dn Known WS=3.03
Boundary for River Rch & Prof#=CornerB,M001            , 4
Up Type= 0
Dn Type= 1
Dn Known WS=2.85
Boundary for River Rch & Prof#=CornerB,M001            , 5
Up Type= 0
Dn Type= 1
Dn Known WS=2.85
Boundary for River Rch & Prof#=CornerB,M001            , 6
Up Type= 0
Dn Type= 1
Dn Known WS=3.03
Boundary for River Rch & Prof#=CornerB,M001            , 7
Up Type= 0
Dn Type= 1
Dn Known WS=3.03
Boundary for River Rch & Prof#=CornerB,M001            , 8
Up Type= 0
Dn Type= 1
Dn Known WS=3.36
Boundary for River Rch & Prof#=CornerB,M001            , 9
Up Type= 0
Dn Type= 1
Dn Known WS=3.36
Boundary for River Rch & Prof#=CornerB,M001            , 10
Up Type= 0
Dn Type= 1
Dn Known WS=2.85
Boundary for River Rch & Prof#=CornerB,M001            , 11
Up Type= 0
Dn Type= 1
Dn Known WS=2.85
Boundary for River Rch & Prof#=CornerB,M001            , 12
Up Type= 0
Dn Type= 1
Dn Known WS=3.03
Boundary for River Rch & Prof#=CornerB,M001            , 13
Up Type= 0
Dn Type= 1
Dn Known WS=3.03
Boundary for River Rch & Prof#=CornerB,M001            , 14
Up Type= 0
Dn Type= 1
Dn Known WS=3.36
Boundary for River Rch & Prof#=CornerB,M001            , 15
Up Type= 0
Dn Type= 1
Dn Known WS=3.36
Boundary for River Rch & Prof#=CornerB,M001            , 16
Up Type= 0
Dn Type= 1
Dn Known WS=2.85
Boundary for River Rch & Prof#=CornerB,M001            , 17
Up Type= 0
Dn Type= 1
Dn Known WS=2.85
Boundary for River Rch & Prof#=CornerB,M001            , 18
Up Type= 0
Dn Type= 1
Dn Known WS=3.03
Boundary for River Rch & Prof#=CornerB,M001            , 19
Up Type= 0
Dn Type= 1
Dn Known WS=3.03
Boundary for River Rch & Prof#=CornerB,M001            , 20
Up Type= 0
Dn Type= 1
Dn Known WS=3.36
Boundary for River Rch & Prof#=CornerB,M001            , 21
Up Type= 0
Dn Type= 1
Dn Known WS=3.36
Gate Openings=CornerB         ,M003            ,2263.0  ,Gate #1     ,
       0       0       0       0       0       0       0       0       0       0
       0       0       0       0       0       0       0       0       0       0
       0       0       0       0       0       0       0       0       0       0
       0       0       0       0       0       0       0       0       0       0
   2.134       0   2.134       0   2.134       0   2.134       0       0       0
DSS Import GetInterval= 0
DSS Import GetPeak= 0
DSS Import FillOption= 0

--- Corner_Brook2.f02 (steady flow) ---

Flow Title=100yr
Program Version=4.10
Number of Profiles= 21
Profile Names=100Year-Existing,AMEC-100yr-2020-90%,AMEC-100yr-2020-Max,AMEC-100yr-2050-90%,AMEC-100yr-2050-Max,AMEC-100yr-2080-90%,AMEC-100yr-2080-Max,FINIIS-100yr-2050-90%,FINIIS-100yr-2050-Max,CGCM2-100yr-2020-90%,CGCM2-100yr-2020-Max,CGCM2-100yr-2050-90%,CGCM2-100yr-2050-Max,CGCM2-100yr-2080-90%,CGCM2-100yr-2080-Max,HADCM3-100yr-2020-90%,HADCM3-100yr-2020-Max,HADCM3-100yr-2050-90%,HADCM3-100yr-2050-Max,HADCM3-100yr-2080-90%,HADCM3-100yr-2080-Max
River Rch & RM=BellsB,TR001           ,178.13
    17.7    19.1    19.8    19.4    20.1    20.3    21.4    42.4    41.7    29.4
    28.9    30.1    29.5    35.4    36.3    24.4    23.9      41    40.3    27.6
    28.2
River Rch & RM=BellsB,M002            ,5166.11
    14.6    15.7    16.2    15.9    16.4    16.7    17.4      34    33.4    23.8
    23.4    24.4    23.9    28.6    29.2    19.9    19.5    32.9    32.3    22.4
    22.9
River Rch & RM=BellsB,M002            ,4436.28
    26.5    28.4    29.3    28.8    29.7    30.1    31.1    59.4    59.7    42.4
    41.6    43.4    42.6    50.9      52    35.2    34.6    58.8    57.7    39.7
    40.6
River Rch & RM=BellsB,M002            ,3329.08
    33.4    35.9    37.1    36.4    37.6    38.1    39.9    73.6    75.2    52.8
    51.9    54.1    53.1    63.9    65.3    44.2    43.5    74.1    72.7    49.5
    50.6
River Rch & RM=BellsB,M002            ,2295.83
    35.9    38.7    39.9    39.2    40.5    41.1    43.1    78.6      81    56.6
    55.6      58    56.9    68.6    70.2    48.2    47.5    79.7    78.2    52.9
    54.2
River Rch & RM=BellsB,M001            ,1582.05
    57.2    61.6    63.7    62.5    64.6    65.5    68.8   126.8   130.2    90.9
    89.3    93.1    91.4   110.3     113      78    76.7   128.1   125.8    85.3
    87.2
River Rch & RM=BellsB,M001            ,816.09
    58.5    63.1    65.2      64    66.2    67.1    70.5   129.2   133.2    92.9
    91.3    95.1    93.4   112.8   115.6    79.9    78.7     131   128.6    87.5
    89.4
River Rch & RM=CornerB,M004            ,2888.71
   187.3   204.1   212.4   207.1   215.6   217.5   227.5   453.2   448.3     314
   310.6   321.4   317.9   379.6   387.2   260.1   257.3   438.1   433.4   294.8
   300.8
River Rch & RM=CornerB,TR001           ,206.04
    32.1    34.8      36    35.3    36.6      37    38.8    76.7    75.6    53.2
    52.5    54.5    53.7    64.2    65.8    44.2    43.6    74.2    73.1      50
    51.2
River Rch & RM=CornerB,M003            ,2689.92
   205.2     224   233.3   227.2   236.7   238.9     250   503.2   497.7   346.6
   342.8   354.9   351.1   420.2   428.8   286.3   283.3   486.2   480.8   325.2
   331.9
River Rch & RM=CornerB,M003            ,2267.71
   205.6   224.5   233.7   227.7   237.2   239.4   250.4     504   498.6   347.2
   343.5   355.5   351.7   420.9   429.5   286.8   283.8     487   481.7   325.8
   332.4
River Rch & RM=CornerB,TR002           ,21.04
    12.2    13.1    13.5    13.3    13.7    13.9    14.5    28.1    27.6    19.8
    19.4    20.2    19.8    23.6    24.1    16.5    16.2    27.2    26.7    18.6
      19
River Rch & RM=CornerB,M002            ,1826.39
   207.6   226.7   236.1     230   239.6   241.7   252.9   509.2   503.7   350.7
     347   359.1   355.3   425.2   433.8   289.7   286.7     492   486.7     329
   335.8
River Rch & RM=CornerB,M002            ,1539.91
   206.4   225.5     235   228.8   238.5   240.6   251.8   508.8   503.4   349.7
     346   358.1   354.3   424.8   433.3   288.6   285.6   491.6   486.4     328
   334.6
River Rch & RM=CornerB,M002            ,915.75
   205.5   224.7   234.1     228   237.7   239.7   250.9   508.6   503.2     349
   345.4   357.4   353.7   424.3   432.8   287.9   284.9   491.3   486.1   327.3
   333.9
River Rch & RM=CornerB,M002            ,828.33
   199.7   218.7   228.1   221.9   231.6   233.6   244.6   500.9   495.7   341.9
   338.4   350.4   346.7   416.8   425.1   281.3   278.4   483.6   478.6   320.4
   326.8
River Rch & RM=CornerB,M001            ,659.37
   209.9   230.3   240.4   233.7   244.1     246   257.5   529.8   524.4   360.8
   357.3   369.7   366.1   440.4   448.9   296.6   293.7   511.4   506.3   337.9
   344.5
Boundary for River Rch & Prof#=BellsB,TR001           , 1
Up Type= 3
Up Slope=0.043
Dn Type= 0
Boundary for River Rch & Prof#=BellsB,TR001           , 2
Up Type= 3
Up Slope=0.043
Dn Type= 0
Boundary for River Rch & Prof#=BellsB,TR001           , 3
Up Type= 3
Up Slope=0.043
Dn Type= 0
Boundary for River Rch & Prof#=BellsB,TR001           , 4
Up Type= 3
Up Slope=0.043
Dn Type= 0
Boundary for River Rch & Prof#=BellsB,TR001           , 5
Up Type= 3
Up Slope=0.043
Dn Type= 0
Boundary for River Rch & Prof#=BellsB,TR001           , 6
Up Type= 3
Up Slope=0.043
Dn Type= 0
Boundary for River Rch & Prof#=BellsB,TR001           , 7
Up Type= 3
Up Slope=0.043
Dn Type= 0
Boundary for River Rch & Prof#=BellsB,TR001           , 8
Up Type= 3
Up Slope=0.043
Dn Type= 0
Boundary for River Rch & Prof#=BellsB,TR001           , 9
Up Type= 3
Up Slope=0.043
Dn Type= 0
Boundary for River Rch & Prof#=BellsB,TR001           , 10
Up Type= 3
Up Slope=0.043
Dn Type= 0
Boundary for River Rch & Prof#=BellsB,TR001           , 11
Up Type= 3
Up Slope=0.043
Dn Type= 0
Boundary for River Rch & Prof#=BellsB,TR001           , 12
Up Type= 3
Up Slope=0.043
Dn Type= 0
Boundary for River Rch & Prof#=BellsB,TR001           , 13
Up Type= 3
Up Slope=0.043
Dn Type= 0
Boundary for River Rch & Prof#=BellsB,TR001           , 14
Up Type= 3
Up Slope=0.043
Dn Type= 0
Boundary for River Rch & Prof#=BellsB,TR001           , 15
Up Type= 3
Up Slope=0.043
Dn Type= 0
Boundary for River Rch & Prof#=BellsB,TR001           , 16
Up Type= 3
Up Slope=0.043
Dn Type= 0
Boundary for River Rch & Prof#=BellsB,TR001           , 17
Up Type= 3
Up Slope=0.043
Dn Type= 0
Boundary for River Rch & Prof#=BellsB,TR001           , 18
Up Type= 3
Up Slope=0.043
Dn Type= 0
Boundary for River Rch & Prof#=BellsB,TR001           , 19
Up Type= 3
Up Slope=0.043
Dn Type= 0
Boundary for River Rch & Prof#=BellsB,TR001           , 20
Up Type= 3
Up Slope=0.043
Dn Type= 0
Boundary for River Rch & Prof#=BellsB,TR001           , 21
Up Type= 3
Up Slope=0.043
Dn Type= 0
Boundary for River Rch & Prof#=BellsB,M002            , 1
Up Type= 3
Up Slope=0.013
Dn Type= 0
Boundary for River Rch & Prof#=BellsB,M002            , 2
Up Type= 3
Up Slope=0.013
Dn Type= 0
Boundary for River Rch & Prof#=BellsB,M002            , 3
Up Type= 3
Up Slope=0.013
Dn Type= 0
Boundary for River Rch & Prof#=BellsB,M002            , 4
Up Type= 3
Up Slope=0.013
Dn Type= 0
Boundary for River Rch & Prof#=BellsB,M002            , 5
Up Type= 3
Up Slope=0.013
Dn Type= 0
Boundary for River Rch & Prof#=BellsB,M002            , 6
Up Type= 3
Up Slope=0.013
Dn Type= 0
Boundary for River Rch & Prof#=BellsB,M002            , 7
Up Type= 3
Up Slope=0.013
Dn Type= 0
Boundary for River Rch & Prof#=BellsB,M002            , 8
Up Type= 3
Up Slope=0.013
Dn Type= 0
Boundary for River Rch & Prof#=BellsB,M002            , 9
Up Type= 3
Up Slope=0.013
Dn Type= 0
Boundary for River Rch & Prof#=BellsB,M002            , 10
Up Type= 3
Up Slope=0.013
Dn Type= 0
Boundary for River Rch & Prof#=BellsB,M002            , 11
Up Type= 3
Up Slope=0.013
Dn Type= 0
Boundary for River Rch & Prof#=BellsB,M002            , 12
Up Type= 3
Up Slope=0.013
Dn Type= 0
Boundary for River Rch & Prof#=BellsB,M002            , 13
Up Type= 3
Up Slope=0.013
Dn Type= 0
Boundary for River Rch & Prof#=BellsB,M002            , 14
Up Type= 3
Up Slope=0.013
Dn Type= 0
Boundary for River Rch & Prof#=BellsB,M002            , 15
Up Type= 3
Up Slope=0.013
Dn Type= 0
Boundary for River Rch & Prof#=BellsB,M002            , 16
Up Type= 3
Up Slope=0.013
Dn Type= 0
Boundary for River Rch & Prof#=BellsB,M002            , 17
Up Type= 3
Up Slope=0.013
Dn Type= 0
Boundary for River Rch & Prof#=BellsB,M002            , 18
Up Type= 3
Up Slope=0.013
Dn Type= 0
Boundary for River Rch & Prof#=BellsB,M002            , 19
Up Type= 3
Up Slope=0.013
Dn Type= 0
Boundary for River Rch & Prof#=BellsB,M002            , 20
Up Type= 3
Up Slope=0.013
Dn Type= 0
Boundary for River Rch & Prof#=BellsB,M002            , 21
Up Type= 3
Up Slope=0.013
Dn Type= 0
Boundary for River Rch & Prof#=BellsB,M001            , 1
Up Type= 0
Dn Type= 0
Boundary for River Rch & Prof#=BellsB,M001            , 2
Up Type= 0
Dn Type= 0
Boundary for River Rch & Prof#=BellsB,M001            , 3
Up Type= 0
Dn Type= 0
Boundary for River Rch & Prof#=BellsB,M001            , 4
Up Type= 0
Dn Type= 0
Boundary for River Rch & Prof#=BellsB,M001            , 5
Up Type= 0
Dn Type= 0
Boundary for River Rch & Prof#=BellsB,M001            , 6
Up Type= 0
Dn Type= 0
Boundary for River Rch & Prof#=BellsB,M001            , 7
Up Type= 0
Dn Type= 0
Boundary for River Rch & Prof#=BellsB,M001            , 8
Up Type= 0
Dn Type= 0
Boundary for River Rch & Prof#=BellsB,M001            , 9
Up Type= 0
Dn Type= 0
Boundary for River Rch & Prof#=BellsB,M001            , 10
Up Type= 0
Dn Type= 0
Boundary for River Rch & Prof#=BellsB,M001            , 11
Up Type= 0
Dn Type= 0
Boundary for River Rch & Prof#=BellsB,M001            , 12
Up Type= 0
Dn Type= 0
Boundary for River Rch & Prof#=BellsB,M001            , 13
Up Type= 0
Dn Type= 0
Boundary for River Rch & Prof#=BellsB,M001            , 14
Up Type= 0
Dn Type= 0
Boundary for River Rch & Prof#=BellsB,M001            , 15
Up Type= 0
Dn Type= 0
Boundary for River Rch & Prof#=BellsB,M001            , 16
Up Type= 0
Dn Type= 0
Boundary for River Rch & Prof#=BellsB,M001            , 17
Up Type= 0
Dn Type= 0
Boundary for River Rch & Prof#=BellsB,M001            , 18
Up Type= 0
Dn Type= 0
Boundary for River Rch & Prof#=BellsB,M001            , 19
Up Type= 0
Dn Type= 0
Boundary for River Rch & Prof#=BellsB,M001            , 20
Up Type= 0
Dn Type= 0
Boundary for River Rch & Prof#=BellsB,M001            , 21
Up Type= 0
Dn Type= 0
Boundary for River Rch & Prof#=CornerB,M004            , 1
Up Type= 3
Up Slope=0.006
Dn Type= 0
Boundary for River Rch & Prof#=CornerB,M004            , 2
Up Type= 3
Up Slope=0.006
Dn Type= 0
Boundary for River Rch & Prof#=CornerB,M004            , 3
Up Type= 3
Up Slope=0.006
Dn Type= 0
Boundary for River Rch & Prof#=CornerB,M004            , 4
Up Type= 3
Up Slope=0.006
Dn Type= 0
Boundary for River Rch & Prof#=CornerB,M004            , 5
Up Type= 3
Up Slope=0.006
Dn Type= 0
Boundary for River Rch & Prof#=CornerB,M004            , 6
Up Type= 3
Up Slope=0.006
Dn Type= 0
Boundary for River Rch & Prof#=CornerB,M004            , 7
Up Type= 3
Up Slope=0.006
Dn Type= 0
Boundary for River Rch & Prof#=CornerB,M004            , 8
Up Type= 3
Up Slope=0.006
Dn Type= 0
Boundary for River Rch & Prof#=CornerB,M004            , 9
Up Type= 3
Up Slope=0.006
Dn Type= 0
Boundary for River Rch & Prof#=CornerB,M004            , 10
Up Type= 3
Up Slope=0.006
Dn Type= 0
Boundary for River Rch & Prof#=CornerB,M004            , 11
Up Type= 3
Up Slope=0.006
Dn Type= 0
Boundary for River Rch & Prof#=CornerB,M004            , 12
Up Type= 3
Up Slope=0.006
Dn Type= 0
Boundary for River Rch & Prof#=CornerB,M004            , 13
Up Type= 3
Up Slope=0.006
Dn Type= 0
Boundary for River Rch & Prof#=CornerB,M004            , 14
Up Type= 3
Up Slope=0.006
Dn Type= 0
Boundary for River Rch & Prof#=CornerB,M004            , 15
Up Type= 3
Up Slope=0.006
Dn Type= 0
Boundary for River Rch & Prof#=CornerB,M004            , 16
Up Type= 3
Up Slope=0.006
Dn Type= 0
Boundary for River Rch & Prof#=CornerB,M004            , 17
Up Type= 3
Up Slope=0.006
Dn Type= 0
Boundary for River Rch & Prof#=CornerB,M004            , 18
Up Type= 3
Up Slope=0.006
Dn Type= 0
Boundary for River Rch & Prof#=CornerB,M004            , 19
Up Type= 3
Up Slope=0.006
Dn Type= 0
Boundary for River Rch & Prof#=CornerB,M004            , 20
Up Type= 3
Up Slope=0.006
Dn Type= 0
Boundary for River Rch & Prof#=CornerB,M004            , 21
Up Type= 3
Up Slope=0.006
Dn Type= 0
Boundary for River Rch & Prof#=CornerB,TR001           , 1
Up Type= 3
Up Slope=0.042
Dn Type= 0
Boundary for River Rch & Prof#=CornerB,TR001           , 2
Up Type= 3
Up Slope=0.042
Dn Type= 0
Boundary for River Rch & Prof#=CornerB,TR001           , 3
Up Type= 3
Up Slope=0.042
Dn Type= 0
Boundary for River Rch & Prof#=CornerB,TR001           , 4
Up Type= 3
Up Slope=0.042
Dn Type= 0
Boundary for River Rch & Prof#=CornerB,TR001           , 5
Up Type= 3
Up Slope=0.042
Dn Type= 0
Boundary for River Rch & Prof#=CornerB,TR001           , 6
Up Type= 3
Up Slope=0.042
Dn Type= 0
Boundary for River Rch & Prof#=CornerB,TR001           , 7
Up Type= 3
Up Slope=0.042
Dn Type= 0
Boundary for River Rch & Prof#=CornerB,TR001           , 8
Up Type= 3
Up Slope=0.042
Dn Type= 0
Boundary for River Rch & Prof#=CornerB,TR001           , 9
Up Type= 3
Up Slope=0.042
Dn Type= 0
Boundary for River Rch & Prof#=CornerB,TR001           , 10
Up Type= 3
Up Slope=0.042
Dn Type= 0
Boundary for River Rch & Prof#=CornerB,TR001           , 11
Up Type= 3
Up Slope=0.042
Dn Type= 0
Boundary for River Rch & Prof#=CornerB,TR001           , 12
Up Type= 3
Up Slope=0.042
Dn Type= 0
Boundary for River Rch & Prof#=CornerB,TR001           , 13
Up Type= 3
Up Slope=0.042
Dn Type= 0
Boundary for River Rch & Prof#=CornerB,TR001           , 14
Up Type= 3
Up Slope=0.042
Dn Type= 0
Boundary for River Rch & Prof#=CornerB,TR001           , 15
Up Type= 3
Up Slope=0.042
Dn Type= 0
Boundary for River Rch & Prof#=CornerB,TR001           , 16
Up Type= 3
Up Slope=0.042
Dn Type= 0
Boundary for River Rch & Prof#=CornerB,TR001           , 17
Up Type= 3
Up Slope=0.042
Dn Type= 0
Boundary for River Rch & Prof#=CornerB,TR001           , 18
Up Type= 3
Up Slope=0.042
Dn Type= 0
Boundary for River Rch & Prof#=CornerB,TR001           , 19
Up Type= 3
Up Slope=0.042
Dn Type= 0
Boundary for River Rch & Prof#=CornerB,TR001           , 20
Up Type= 3
Up Slope=0.042
Dn Type= 0
Boundary for River Rch & Prof#=CornerB,TR001           , 21
Up Type= 3
Up Slope=0.042
Dn Type= 0
Boundary for River Rch & Prof#=CornerB,M003            , 1
Up Type= 0
Dn Type= 0
Boundary for River Rch & Prof#=CornerB,M003            , 2
Up Type= 0
Dn Type= 0
Boundary for River Rch & Prof#=CornerB,M003            , 3
Up Type= 0
Dn Type= 0
Boundary for River Rch & Prof#=CornerB,M003            , 4
Up Type= 0
Dn Type= 0
Boundary for River Rch & Prof#=CornerB,M003            , 5
Up Type= 0
Dn Type= 0
Boundary for River Rch & Prof#=CornerB,M003            , 6
Up Type= 0
Dn Type= 0
Boundary for River Rch & Prof#=CornerB,M003            , 7
Up Type= 0
Dn Type= 0
Boundary for River Rch & Prof#=CornerB,M003            , 8
Up Type= 0
Dn Type= 0
Boundary for River Rch & Prof#=CornerB,M003            , 9
Up Type= 0
Dn Type= 0
Boundary for River Rch & Prof#=CornerB,M003            , 10
Up Type= 0
Dn Type= 0
Boundary for River Rch & Prof#=CornerB,M003            , 11
Up Type= 0
Dn Type= 0
Boundary for River Rch & Prof#=CornerB,M003            , 12
Up Type= 0
Dn Type= 0
Boundary for River Rch & Prof#=CornerB,M003            , 13
Up Type= 0
Dn Type= 0
Boundary for River Rch & Prof#=CornerB,M003            , 14
Up Type= 0
Dn Type= 0
Boundary for River Rch & Prof#=CornerB,M003            , 15
Up Type= 0
Dn Type= 0
Boundary for River Rch & Prof#=CornerB,M003            , 16
Up Type= 0
Dn Type= 0
Boundary for River Rch & Prof#=CornerB,M003            , 17
Up Type= 0
Dn Type= 0
Boundary for River Rch & Prof#=CornerB,M003            , 18
Up Type= 0
Dn Type= 0
Boundary for River Rch & Prof#=CornerB,M003            , 19
Up Type= 0
Dn Type= 0
Boundary for River Rch & Prof#=CornerB,M003            , 20
Up Type= 0
Dn Type= 0
Boundary for River Rch & Prof#=CornerB,M003            , 21
Up Type= 0
Dn Type= 0
Boundary for River Rch & Prof#=CornerB,TR002           , 1
Up Type= 3
Up Slope=0.15
Dn Type= 0
Boundary for River Rch & Prof#=CornerB,TR002           , 2
Up Type= 3
Up Slope=0.15
Dn Type= 0
Boundary for River Rch & Prof#=CornerB,TR002           , 3
Up Type= 3
Up Slope=0.15
Dn Type= 0
Boundary for River Rch & Prof#=CornerB,TR002           , 4
Up Type= 3
Up Slope=0.15
Dn Type= 0
Boundary for River Rch & Prof#=CornerB,TR002           , 5
Up Type= 3
Up Slope=0.15
Dn Type= 0
Boundary for River Rch & Prof#=CornerB,TR002           , 6
Up Type= 3
Up Slope=0.15
Dn Type= 0
Boundary for River Rch & Prof#=CornerB,TR002           , 7
Up Type= 3
Up Slope=0.15
Dn Type= 0
Boundary for River Rch & Prof#=CornerB,TR002           , 8
Up Type= 3
Up Slope=0.15
Dn Type= 0
Boundary for River Rch & Prof#=CornerB,TR002           , 9
Up Type= 3
Up Slope=0.15
Dn Type= 0
Boundary for River Rch & Prof#=CornerB,TR002           , 10
Up Type= 3
Up Slope=0.15
Dn Type= 0
Boundary for River Rch & Prof#=CornerB,TR002           , 11
Up Type= 3
Up Slope=0.15
Dn Type= 0
Boundary for River Rch & Prof#=CornerB,TR002           , 12
Up Type= 3
Up Slope=0.15
Dn Type= 0
Boundary for River Rch & Prof#=CornerB,TR002           , 13
Up Type= 3
Up Slope=0.15
Dn Type= 0
Boundary for River Rch & Prof#=CornerB,TR002           , 14
Up Type= 3
Up Slope=0.15
Dn Type= 0
Boundary for River Rch & Prof#=CornerB,TR002           , 15
Up Type= 3
Up Slope=0.15
Dn Type= 0
Boundary for River Rch & Prof#=CornerB,TR002           , 16
Up Type= 3
Up Slope=0.15
Dn Type= 0
Boundary for River Rch & Prof#=CornerB,TR002           , 17
Up Type= 3
Up Slope=0.15
Dn Type= 0
Boundary for River Rch & Prof#=CornerB,TR002           , 18
Up Type= 3
Up Slope=0.15
Dn Type= 0
Boundary for River Rch & Prof#=CornerB,TR002           , 19
Up Type= 3
Up Slope=0.15
Dn Type= 0
Boundary for River Rch & Prof#=CornerB,TR002           , 20
Up Type= 3
Up Slope=0.15
Dn Type= 0
Boundary for River Rch & Prof#=CornerB,TR002           , 21
Up Type= 3
Up Slope=0.15
Dn Type= 0
Boundary for River Rch & Prof#=CornerB,M002            , 1
Up Type= 0
Dn Type= 0
Boundary for River Rch & Prof#=CornerB,M002            , 2
Up Type= 0
Dn Type= 0
Boundary for River Rch & Prof#=CornerB,M002            , 3
Up Type= 0
Dn Type= 0
Boundary for River Rch & Prof#=CornerB,M002            , 4
Up Type= 0
Dn Type= 0
Boundary for River Rch & Prof#=CornerB,M002            , 5
Up Type= 0
Dn Type= 0
Boundary for River Rch & Prof#=CornerB,M002            , 6
Up Type= 0
Dn Type= 0
Boundary for River Rch & Prof#=CornerB,M002            , 7
Up Type= 0
Dn Type= 0
Boundary for River Rch & Prof#=CornerB,M002            , 8
Up Type= 0
Dn Type= 0
Boundary for River Rch & Prof#=CornerB,M002            , 9
Up Type= 0
Dn Type= 0
Boundary for River Rch & Prof#=CornerB,M002            , 10
Up Type= 0
Dn Type= 0
Boundary for River Rch & Prof#=CornerB,M002            , 11
Up Type= 0
Dn Type= 0
Boundary for River Rch & Prof#=CornerB,M002            , 12
Up Type= 0
Dn Type= 0
Boundary for River Rch & Prof#=CornerB,M002            , 13
Up Type= 0
Dn Type= 0
Boundary for River Rch & Prof#=CornerB,M002            , 14
Up Type= 0
Dn Type= 0
Boundary for River Rch & Prof#=CornerB,M002            , 15
Up Type= 0
Dn Type= 0
Boundary for River Rch & Prof#=CornerB,M002            , 16
Up Type= 0
Dn Type= 0
Boundary for River Rch & Prof#=CornerB,M002            , 17
Up Type= 0
Dn Type= 0
Boundary for River Rch & Prof#=CornerB,M002            , 18
Up Type= 0
Dn Type= 0
Boundary for River Rch & Prof#=CornerB,M002            , 19
Up Type= 0
Dn Type= 0
Boundary for River Rch & Prof#=CornerB,M002            , 20
Up Type= 0
Dn Type= 0
Boundary for River Rch & Prof#=CornerB,M002            , 21
Up Type= 0
Dn Type= 0
Boundary for River Rch & Prof#=CornerB,M001            , 1
Up Type= 0
Dn Type= 1
Dn Known WS=2.8
Boundary for River Rch & Prof#=CornerB,M001            , 2
Up Type= 0
Dn Type= 1
Dn Known WS=2.85
Boundary for River Rch & Prof#=CornerB,M001            , 3
Up Type= 0
Dn Type= 1
Dn Known WS=2.85
Boundary for River Rch & Prof#=CornerB,M001            , 4
Up Type= 0
Dn Type= 1
Dn Known WS=3.03
Boundary for River Rch & Prof#=CornerB,M001            , 5
Up Type= 0
Dn Type= 1
Dn Known WS=3.03
Boundary for River Rch & Prof#=CornerB,M001            , 6
Up Type= 0
Dn Type= 1
Dn Known WS=3.36
Boundary for River Rch & Prof#=CornerB,M001            , 7
Up Type= 0
Dn Type= 1
Dn Known WS=3.36
Boundary for River Rch & Prof#=CornerB,M001            , 8
Up Type= 0
Dn Type= 1
Dn Known WS=3.03
Boundary for River Rch & Prof#=CornerB,M001            , 9
Up Type= 0
Dn Type= 1
Dn Known WS=3.03
Boundary for River Rch & Prof#=CornerB,M001            , 10
Up Type= 0
Dn Type= 1
Dn Known WS=2.85
Boundary for River Rch & Prof#=CornerB,M001            , 11
Up Type= 0
Dn Type= 1
Dn Known WS=2.85
Boundary for River Rch & Prof#=CornerB,M001            , 12
Up Type= 0
Dn Type= 1
Dn Known WS=3.03
Boundary for River Rch & Prof#=CornerB,M001            , 13
Up Type= 0
Dn Type= 1
Dn Known WS=3.03
Boundary for River Rch & Prof#=CornerB,M001            , 14
Up Type= 0
Dn Type= 1
Dn Known WS=3.36
Boundary for River Rch & Prof#=CornerB,M001            , 15
Up Type= 0
Dn Type= 1
Dn Known WS=3.36
Boundary for River Rch & Prof#=CornerB,M001            , 16
Up Type= 0
Dn Type= 1
Dn Known WS=2.85
Boundary for River Rch & Prof#=CornerB,M001            , 17
Up Type= 0
Dn Type= 1
Dn Known WS=2.85
Boundary for River Rch & Prof#=CornerB,M001            , 18
Up Type= 0
Dn Type= 1
Dn Known WS=3.03
Boundary for River Rch & Prof#=CornerB,M001            , 19
Up Type= 0
Dn Type= 1
Dn Known WS=3.03
Boundary for River Rch & Prof#=CornerB,M001            , 20
Up Type= 0
Dn Type= 1
Dn Known WS=3.36
Boundary for River Rch & Prof#=CornerB,M001            , 21
Up Type= 0
Dn Type= 1
Dn Known WS=3.36
Gate Openings=CornerB         ,M003            ,2263.0  ,Gate #1     ,
   2.134       0   2.134       0   2.134       0   2.134       0   2.134       0
   2.134       0   2.134       0   2.134       0   2.134       0   2.134       0
   2.134       0   2.134       0   2.134       0   2.134       0   2.134       0
   2.134       0   2.134       0   2.134       0   2.134       0   2.134       0
   2.134       0
DSS Import GetInterval= 0
DSS Import GetPeak= 0
DSS Import FillOption= 0
