HEC-RAS study Corner_Brook2.prj: Corner_Brook2

--- Corner_Brook2.f03 (steady flow) ---

Flow Title=100yr-2013
Program Version=4.10
Number of Profiles= 5
Profile Names=100-Existing,AMEC-100-2020-Max,AMEC-100-2050-Max,FINNIS-100-2050-Max,AMEC-100-2080-Max
River Rch & RM=BellsB,TR001           ,178.13
    17.7    19.8    20.1    41.7    21.4
River Rch & RM=BellsB,M002            ,5166.11
    14.6    16.2    16.4    33.4    17.4
River Rch & RM=BellsB,M002            ,4436.28
    26.5    29.3    29.7    59.7    31.1
River Rch & RM=BellsB,M002            ,3329.08
    33.4    37.1    37.6    75.2    39.9
River Rch & RM=BellsB,M002            ,2295.83
    35.9    39.9    40.5      81    43.1
River Rch & RM=BellsB,M001            ,1582.05
    57.2    63.7    64.6   130.2    68.8
River Rch & RM=BellsB,M001            ,816.09
    58.5    65.2    66.2   133.2    70.5
River Rch & RM=CornerB,M004            ,2888.71
   178.7   201.5   203.8   422.4   215.4
River Rch & RM=CornerB,TR001           ,206.04
    32.1      36    36.6    75.6    38.8
River Rch & RM=CornerB,M003            ,2689.92
   196.3   222.8   225.2   471.5   237.4
River Rch & RM=CornerB,M003            ,2267.71
   196.6   223.3   225.7   472.6   237.9
River Rch & RM=CornerB,TR002           ,21.04
    12.2    13.5    13.7    27.6    14.5
River Rch & RM=CornerB,M002            ,1826.39
   198.6   225.8   228.2   477.8   240.3
River Rch & RM=CornerB,M002            ,1539.91
   197.5   224.6   227.2   477.9   238.9
River Rch & RM=CornerB,M002            ,915.75
   196.6   223.8   226.4   477.9     238
River Rch & RM=CornerB,M002            ,828.33
   190.8   217.9   220.4   470.5   231.8
River Rch & RM=CornerB,M001            ,659.37
     201   230.7   233.5     500   244.9
Boundary for River Rch & Prof#=BellsB,TR001           , 1
Up Type= 3
Up Slope=0.043
Dn Type= 0
Boundary for River Rch & Prof#=BellsB,TR001           , 2
Up Type= 3
Up Slope=0.043
Dn Type= 0
Boundary for River Rch & Prof#=BellsB,TR001           , 3
Up Type= 3
Up Slope=0.043
Dn Type= 0
Boundary for River Rch & Prof#=BellsB,TR001           , 4
Up Type= 3
Up Slope=0.043
Dn Type= 0
Boundary for River Rch & Prof#=BellsB,TR001           , 5
Up Type= 3
Up Slope=0.043
Dn Type= 0
Boundary for River Rch & Prof#=BellsB,M002            , 1
Up Type= 3
Up Slope=0.013
Dn Type= 0
Boundary for River Rch & Prof#=BellsB,M002            , 2
Up Type= 3
Up Slope=0.013
Dn Type= 0
Boundary for River Rch & Prof#=BellsB,M002            , 3
Up Type= 3
Up Slope=0.013
Dn Type= 0
Boundary for River Rch & Prof#=BellsB,M002            , 4
Up Type= 3
Up Slope=0.013
Dn Type= 0
Boundary for River Rch & Prof#=BellsB,M002            , 5
Up Type= 3
Up Slope=0.013
Dn Type= 0
Boundary for River Rch & Prof#=BellsB,M001            , 1
Up Type= 0
Dn Type= 0
Boundary for River Rch & Prof#=BellsB,M001            , 2
Up Type= 0
Dn Type= 0
Boundary for River Rch & Prof#=BellsB,M001            , 3
Up Type= 0
Dn Type= 0
Boundary for River Rch & Prof#=BellsB,M001            , 4
Up Type= 0
Dn Type= 0
Boundary for River Rch & Prof#=BellsB,M001            , 5
Up Type= 0
Dn Type= 0
Boundary for River Rch & Prof#=CornerB,M004            , 1
Up Type= 3
Up Slope=0.006
Dn Type= 0
Boundary for River Rch & Prof#=CornerB,M004            , 2
Up Type= 3
Up Slope=0.006
Dn Type= 0
Boundary for River Rch & Prof#=CornerB,M004            , 3
Up Type= 3
Up Slope=0.006
Dn Type= 0
Boundary for River Rch & Prof#=CornerB,M004            , 4
Up Type= 3
Up Slope=0.006
Dn Type= 0
Boundary for River Rch & Prof#=CornerB,M004            , 5
Up Type= 3
Up Slope=0.006
Dn Type= 0
Boundary for River Rch & Prof#=CornerB,TR001           , 1
Up Type= 3
Up Slope=0.042
Dn Type= 0
Boundary for River Rch & Prof#=CornerB,TR001           , 2
Up Type= 3
Up Slope=0.042
Dn Type= 0
Boundary for River Rch & Prof#=CornerB,TR001           , 3
Up Type= 3
Up Slope=0.042
Dn Type= 0
Boundary for River Rch & Prof#=CornerB,TR001           , 4
Up Type= 3
Up Slope=0.042
Dn Type= 0
Boundary for River Rch & Prof#=CornerB,TR001           , 5
Up Type= 3
Up Slope=0.042
Dn Type= 0
Boundary for River Rch & Prof#=CornerB,M003            , 1
Up Type= 0
Dn Type= 0
Boundary for River Rch & Prof#=CornerB,M003            , 2
Up Type= 0
Dn Type= 0
Boundary for River Rch & Prof#=CornerB,M003            , 3
Up Type= 0
Dn Type= 0
Boundary for River Rch & Prof#=CornerB,M003            , 4
Up Type= 0
Dn Type= 0
Boundary for River Rch & Prof#=CornerB,M003            , 5
Up Type= 0
Dn Type= 0
Boundary for River Rch & Prof#=CornerB,TR002           , 1
Up Type= 3
Up Slope=0.15
Dn Type= 0
Boundary for River Rch & Prof#=CornerB,TR002           , 2
Up Type= 3
Up Slope=0.15
Dn Type= 0
Boundary for River Rch & Prof#=CornerB,TR002           , 3
Up Type= 3
Up Slope=0.15
Dn Type= 0
Boundary for River Rch & Prof#=CornerB,TR002           , 4
Up Type= 3
Up Slope=0.15
Dn Type= 0
Boundary for River Rch & Prof#=CornerB,TR002           , 5
Up Type= 3
Up Slope=0.15
Dn Type= 0
Boundary for River Rch & Prof#=CornerB,M002            , 1
Up Type= 0
Dn Type= 0
Boundary for River Rch & Prof#=CornerB,M002            , 2
Up Type= 0
Dn Type= 0
Boundary for River Rch & Prof#=CornerB,M002            , 3
Up Type= 0
Dn Type= 0
Boundary for River Rch & Prof#=CornerB,M002            , 4
Up Type= 0
Dn Type= 0
Boundary for River Rch & Prof#=CornerB,M002            , 5
Up Type= 0
Dn Type= 0
Boundary for River Rch & Prof#=CornerB,M001            , 1
Up Type= 0
Dn Type= 1
Dn Known WS=2.8
Boundary for River Rch & Prof#=CornerB,M001            , 2
Up Type= 0
Dn Type= 1
Dn Known WS=2.85
Boundary for River Rch & Prof#=CornerB,M001            , 3
Up Type= 0
Dn Type= 1
Dn Known WS=3.03
Boundary for River Rch & Prof#=CornerB,M001            , 4
Up Type= 0
Dn Type= 1
Dn Known WS=3.03
Boundary for River Rch & Prof#=CornerB,M001            , 5
Up Type= 0
Dn Type= 1
Dn Known WS=3.36
Gate Openings=CornerB         ,M003            ,2263.0  ,Gate #1     ,
   2.134       0   2.134       0   2.134       0   2.134       0   2.134       0
DSS Import GetInterval= 0
DSS Import GetPeak= 0
DSS Import FillOption= 0

--- Corner_Brook2.f04 (steady flow) ---

Flow Title=20yr-2013
Program Version=4.10
Number of Profiles= 5
Profile Names=20-Existing,AMEC-20-2020-Max,AMEC-20-2050-Max,FINNIS-20-2050-Max,AMEC-20-2080-Max
River Rch & RM=BellsB,TR001           ,178.13
    12.5    14.8      15    28.6      16
River Rch & RM=BellsB,M002            ,5166.11
    10.4    12.2    12.3    23.1    12.2
River Rch & RM=BellsB,M002            ,4436.28
    18.8    21.9    22.2      41    21.9
River Rch & RM=BellsB,M002            ,3329.08
    23.8    27.5      28    51.1    27.5
River Rch & RM=BellsB,M002            ,2295.83
      26    29.6    30.1    54.8    29.6
River Rch & RM=BellsB,M001            ,1582.05
    41.3    47.3      48    88.3    47.3
River Rch & RM=BellsB,M001            ,816.09
    42.5    48.4    49.2    90.4    48.4
River Rch & RM=CornerB,M004            ,2888.71
   127.5   152.9   154.6     294   152.9
River Rch & RM=CornerB,TR001           ,206.04
    22.9    27.3    27.6    52.4    27.3
River Rch & RM=CornerB,M003            ,2689.92
   140.1   168.1     170   326.9   168.1
River Rch & RM=CornerB,M003            ,2267.71
   140.5   168.5   170.4   327.7   168.5
River Rch & RM=CornerB,TR002           ,21.04
     8.7    10.1    10.3    19.1    10.1
River Rch & RM=CornerB,M002            ,1826.39
     142   170.3   172.2   331.5   170.3
River Rch & RM=CornerB,M002            ,1539.91
   141.5   169.6   171.4   331.4   169.6
River Rch & RM=CornerB,M002            ,915.75
   140.7   168.8   170.6     331   168.8
River Rch & RM=CornerB,M002            ,828.33
   135.9   163.8   165.5   324.3   163.8
River Rch & RM=CornerB,M001            ,659.37
   142.9   173.3     175   344.8   173.3
Boundary for River Rch & Prof#=BellsB,TR001           , 1
Up Type= 3
Up Slope=0.043
Dn Type= 0
Boundary for River Rch & Prof#=BellsB,TR001           , 2
Up Type= 3
Up Slope=0.043
Dn Type= 0
Boundary for River Rch & Prof#=BellsB,TR001           , 3
Up Type= 3
Up Slope=0.043
Dn Type= 0
Boundary for River Rch & Prof#=BellsB,TR001           , 4
Up Type= 3
Up Slope=0.043
Dn Type= 0
Boundary for River Rch & Prof#=BellsB,TR001           , 5
Up Type= 3
Up Slope=0.043
Dn Type= 0
Boundary for River Rch & Prof#=BellsB,M002            , 1
Up Type= 3
Up Slope=0.013
Dn Type= 0
Boundary for River Rch & Prof#=BellsB,M002            , 2
Up Type= 3
Up Slope=0.013
Dn Type= 0
Boundary for River Rch & Prof#=BellsB,M002            , 3
Up Type= 3
Up Slope=0.013
Dn Type= 0
Boundary for River Rch & Prof#=BellsB,M002            , 4
Up Type= 3
Up Slope=0.013
Dn Type= 0
Boundary for River Rch & Prof#=BellsB,M002            , 5
Up Type= 3
Up Slope=0.013
Dn Type= 0
Boundary for River Rch & Prof#=BellsB,M001            , 1
Up Type= 0
Dn Type= 0
Boundary for River Rch & Prof#=BellsB,M001            , 2
Up Type= 0
Dn Type= 0
Boundary for River Rch & Prof#=BellsB,M001            , 3
Up Type= 0
Dn Type= 0
Boundary for River Rch & Prof#=BellsB,M001            , 4
Up Type= 0
Dn Type= 0
Boundary for River Rch & Prof#=BellsB,M001            , 5
Up Type= 0
Dn Type= 0
Boundary for River Rch & Prof#=CornerB,M004            , 1
Up Type= 3
Up Slope=0.006
Dn Type= 0
Boundary for River Rch & Prof#=CornerB,M004            , 2
Up Type= 3
Up Slope=0.006
Dn Type= 0
Boundary for River Rch & Prof#=CornerB,M004            , 3
Up Type= 3
Up Slope=0.006
Dn Type= 0
Boundary for River Rch & Prof#=CornerB,M004            , 4
Up Type= 3
Up Slope=0.006
Dn Type= 0
Boundary for River Rch & Prof#=CornerB,M004            , 5
Up Type= 3
Up Slope=0.006
Dn Type= 0
Boundary for River Rch & Prof#=CornerB,TR001           , 1
Up Type= 3
Up Slope=0.042
Dn Type= 0
Boundary for River Rch & Prof#=CornerB,TR001           , 2
Up Type= 3
Up Slope=0.042
Dn Type= 0
Boundary for River Rch & Prof#=CornerB,TR001           , 3
Up Type= 3
Up Slope=0.042
Dn Type= 0
Boundary for River Rch & Prof#=CornerB,TR001           , 4
Up Type= 3
Up Slope=0.042
Dn Type= 0
Boundary for River Rch & Prof#=CornerB,TR001           , 5
Up Type= 3
Up Slope=0.042
Dn Type= 0
Boundary for River Rch & Prof#=CornerB,M003            , 1
Up Type= 0
Dn Type= 0
Boundary for River Rch & Prof#=CornerB,M003            , 2
Up Type= 0
Dn Type= 0
Boundary for River Rch & Prof#=CornerB,M003            , 3
Up Type= 0
Dn Type= 0
Boundary for River Rch & Prof#=CornerB,M003            , 4
Up Type= 0
Dn Type= 0
Boundary for River Rch & Prof#=CornerB,M003            , 5
Up Type= 0
Dn Type= 0
Boundary for River Rch & Prof#=CornerB,TR002           , 1
Up Type= 3
Up Slope=0.15
Dn Type= 0
Boundary for River Rch & Prof#=CornerB,TR002           , 2
Up Type= 3
Up Slope=0.15
Dn Type= 0
Boundary for River Rch & Prof#=CornerB,TR002           , 3
Up Type= 3
Up Slope=0.15
Dn Type= 0
Boundary for River Rch & Prof#=CornerB,TR002           , 4
Up Type= 3
Up Slope=0.15
Dn Type= 0
Boundary for River Rch & Prof#=CornerB,TR002           , 5
Up Type= 3
Up Slope=0.15
Dn Type= 0
Boundary for River Rch & Prof#=CornerB,M002            , 1
Up Type= 0
Dn Type= 0
Boundary for River Rch & Prof#=CornerB,M002            , 2
Up Type= 0
Dn Type= 0
Boundary for River Rch & Prof#=CornerB,M002            , 3
Up Type= 0
Dn Type= 0
Boundary for River Rch & Prof#=CornerB,M002            , 4
Up Type= 0
Dn Type= 0
Boundary for River Rch & Prof#=CornerB,M002            , 5
Up Type= 0
Dn Type= 0
Boundary for River Rch & Prof#=CornerB,M001            , 1
Up Type= 0
Dn Type= 1
Dn Known WS=2.8
Boundary for River Rch & Prof#=CornerB,M001            , 2
Up Type= 0
Dn Type= 1
Dn Known WS=2.85
Boundary for River Rch & Prof#=CornerB,M001            , 3
Up Type= 0
Dn Type= 1
Dn Known WS=3.03
Boundary for River Rch & Prof#=CornerB,M001            , 4
Up Type= 0
Dn Type= 1
Dn Known WS=3.03
Boundary for River Rch & Prof#=CornerB,M001            , 5
Up Type= 0
Dn Type= 1
Dn Known WS=3.36
Gate Openings=CornerB         ,M003            ,2263.0  ,Gate #1     ,
   2.134       0   2.134       0   2.134       0   2.134       0   2.134       0
DSS Import GetInterval= 0
DSS Import GetPeak= 0
DSS Import FillOption= 0

--- Corner_Brook2.g01 (geometry) ---

Geom Title=CB_no_below_waterline
Program Version=4.10
BEGIN GEOM DESCRIPTION:
Created based on a TIN with 1 z tolerance
END GEOM DESCRIPTION:

Junct Name=1
Junct Desc=, 0 , 0 ,-1 ,0
Up River,Reach=CornerB         ,M002
Up River,Reach=BellsB          ,M001
Dn River,Reach=CornerB         ,M001
Junc L&A=29.8,
Junc L&A=20.5,0

Junct Name=3
Junct Desc=, 0 , 0 ,-1 ,0
Up River,Reach=CornerB         ,M003
Up River,Reach=CornerB         ,TR002
Dn River,Reach=CornerB         ,M002
Junc L&A=46.25,
Junc L&A=18.08,0

Junct Name=5
Junct Desc=, 0 , 0 ,-1 ,0
Up River,Reach=CornerB         ,M004
Up River,Reach=CornerB         ,TR001
Dn River,Reach=CornerB         ,M003
Junc L&A=42.09,
Junc L&A=21.3,0

Junct Name=8
Junct Desc=, 0 , 0 ,-1 ,0
Up River,Reach=BellsB          ,M002
Up River,Reach=BellsB          ,TR001
Dn River,Reach=BellsB          ,M001
Junc L&A=6.47,
Junc L&A=12.15,

River Reach=BellsB          ,TR001
Reach XY= 21
344257.073913574 5422744.4309082344255.4655151375422747.44512939
344251.8466796885422749.35412598344246.4182739265422753.37310791
 344240.386718755422759.60247803344234.2293090825422768.79211426
 344229.40411377 5422778.1362915 344227.293090825422782.85852051
344223.7747192385422785.47088623344199.6320800785422823.99731445
344195.6109008795422830.12628174344194.1030883795422839.06848145
344192.3941040045422845.09710693344189.9815063485422849.01568604
344186.3624877935422852.13031006344177.4935302735422855.59729004
344168.0441284185422861.22387695344159.0972900395422868.85992432
344152.8646850595422877.60131836344149.5474853525422883.42871094
344144.2833251955422894.11730957

Type RM Length L Ch R = 1 ,178.13  ,18.25,18.27,18.06
XS GIS Cut Line= 6
344234.4996948245422720.95068359344238.9260864265422731.27270508
344238.0407104495422749.41009521344253.2380981455422758.25750732
344279.2062988285422758.69989014344288.9442749025422755.16088867
#Sta/Elev= 29
       0   100.6    1.07  100.17    1.36   100.1    3.95   99.29    6.84   98.69
   11.23   98.43   26.64   97.18   26.75   97.17   29.39   97.06   29.64   97.06
    33.3   95.27   34.92    94.8    37.4   93.66   38.11   93.33   39.46   93.14
   39.72   93.11   40.89  93.708   43.36   94.97   44.56    95.4   46.98   96.42
    48.3   96.87   49.69   96.98   50.19   97.07   66.89      98   72.95   99.37
    79.9  100.72   80.71  100.84   82.12  100.98   83.31  101.11
#Mann= 3 , 0 , 0
       0    .055       0    37.4    .035       0   40.89    .055       0
Bank Sta=37.4,40.89
XS Rating Curve= 0 ,0
Exp/Cntr=0.3,0.1

Type RM Length L Ch R = 1 ,159.86  ,19.69,20.32,20.7
XS GIS Cut Line= 2
344199.8156738285422748.48608398344269.362304688 5422788.0244751
#Sta/Elev= 25
       0  100.72    5.48   98.62    7.71   97.22   12.75   96.95   16.31   96.67
   22.63   96.54   26.89   96.37   32.21   96.16   32.29   96.14   33.23   95.54
   38.95   92.89      39   92.86   39.61   92.56   40.09   92.35   40.73   92.43
      41   92.46   42.58  92.644   44.18   92.83   45.24   93.38   51.06   96.33
   59.79   96.63    70.5   96.86   73.81   96.97   79.98   98.32      80   98.32
#Mann= 3 , 0 , 0
       0    .055       0   39.61    .035       0   42.58    .055       0
Bank Sta=39.61,42.58
XS Rating Curve= 0 ,0
Exp/Cntr=0.3,0.1

Type RM Length L Ch R = 1 ,139.54  ,49.06,48.13,33.83
XS GIS Cut Line= 5
       344187.04     5422775.179      344200.338      5422782.01
      344217.269     5422780.434      344217.269     5422780.434
      344255.016     5422806.982
#Sta/Elev= 30
       0     100     1.7      99    3.45      98    5.35      97    7.53      96
   10.51      95   14.95      96   24.47      96   26.94   96.28   32.46   96.28
   33.74      96   35.57      95   36.96      94   38.56      93   38.84   93.02
  38.845   92.11   38.85   91.14   38.92   91.14   39.81   91.14   40.26   91.13
    41.3   91.13   41.31   92.11   42.23    92.2   43.18      93   46.09      94
   47.56      95   49.89      96   52.35      97   60.24   97.09    78.1   97.09
#Mann= 3 , 0 , 0
       0    .055       0  38.845    .035       0   41.31    .055       0
#XS Ineff= 2 , 0
   14.95   38.92   96.28   41.32   14.95   96.78
Permanent Ineff=
       F       F
Bank Sta=38.845,41.31
XS Rating Curve= 0 ,0
Exp/Cntr=0.5,0.3

Type RM Length L Ch R = 2 ,100     ,,,
BEGIN DESCRIPTION:
O'Connell Drive/Mount Batten Road (Structure #2130)
END DESCRIPTION:
Bridge Culvert--1,0,-1,-1, 0
Deck Dist Width WeirC Skew NumUp NumDn MinLoCord MaxHiCord MaxSubmerge Is_Ogee
12,19.2,1.67,0, 7, 8, 95, , 0.98, 0, 0.73,0.57,,
   14.95   20.39   39.15   46.73   52.28   66.99    78.1
   95.92   95.85   96.78      97   97.05      97   97.09
                                                        
       0   19.48   28.32   36.51   40.19   45.24   49.91   66.38
      97   95.92   95.85      96      96   95.71   95.42      97
                                                                
BR Coef=-1 , 0 , 0 ,, 0 ,,,0.8,-1,,0,
WSPro=,,,, 1 ,,,, 0 ,,,, 0 ,,,,-1 ,-1 ,-1 , 0 , 0 , 0 , 0 , 0
Culvert=1,2.4,,44.2,0.03,0.7,1,2,2,91.13,40.12,89.49,40.27,Culvert #1  , 0 ,1.4
Culvert Bottom n=0.03
BC Design=,, 0 ,, 0 ,,,,,,
BC Use User HTab Curves=0
BC User HTab FreeFlow(D)= 0

Type RM Length L Ch R = 1 ,91.42   ,3.23,3.25,0.95
XS GIS Cut Line= 6
344176.3275146485422793.74768066344187.5899047855422816.60327148
344192.6146850595422823.52929688344201.1046752935422826.99230957
344212.5405273445422816.77648926344218.2583007815422811.40887451
#Sta/Elev= 19
       0      97   27.82      96    29.8      95   31.53      94   33.34      93
    36.2      92   38.17   91.55   38.37      90   39.17  89.759   40.06   89.49
   40.82   89.49   41.03   89.49   41.29  89.933   41.94   91.04   43.13      91
   46.01      92   49.33      93   52.76      94   66.38      96
#Mann= 3 , 0 , 0
       0    .055       0   38.37    .035       0   41.29    .055       0
#XS Ineff= 2 , 0
       0   39.07   93.65   41.47       0   93.65
Permanent Ineff=
       F       F
Bank Sta=38.37,41.29
XS Rating Curve= 0 ,0
Exp/Cntr=0.5,0.3

Type RM Length L Ch R = 1 ,88.17   ,2.5,4.05,10.03
XS GIS Cut Line= 6
344174.2482910165422796.34509277344185.5106811525422819.20068359
344190.5355224615422826.12652588344199.0255126955422829.58947754
344210.4613037115422819.37371826344216.1790771485422814.00610352
#Sta/Elev= 24
       0   97.07   25.47   96.22   25.48   96.21   34.04   92.08   34.66   91.89
   34.86   91.86   35.62   91.59   36.82   90.72   39.14   89.63   39.42   89.47
   40.45  88.864   40.78   88.67   41.92   88.75   43.21   88.84   44.37    89.1
   47.56   91.21    56.5   94.19   57.23   94.44   57.28   94.45   57.55   94.52
   58.54   94.81   61.75   95.78   63.05   95.86   66.38   95.95
#Mann= 3 , 0 , 0
       0    .055       0   40.45    .035       0   43.21    .055       0
Bank Sta=40.45,43.21
XS Rating Curve= 0 ,0
Exp/Cntr=0.3,0.1

Type RM Length L Ch R = 1 ,84.12   ,3.03,4.98,8.8
XS GIS Cut Line= 6
344172.6889038095422796.34509277344187.4166870125422824.04870605
344193.3076782235422831.49407959344199.372070313 5422834.0914917
344213.0603027345422825.26068115344222.7633056645422817.64227295
#Sta/Elev= 24
       0   97.12   26.05   96.23   31.38   93.56   35.51   91.59   35.77   91.44
    36.2   91.36   36.38   91.33   37.44   91.06    39.2   90.27   40.87   89.28
   41.55   88.88   42.87  88.102   43.28   87.86   44.32   87.93   47.47   88.14
   51.66   89.03   52.72   89.72   55.22   90.47   61.86   94.27   63.76   94.37
   68.59   94.62    71.2   95.37   71.88   95.41   76.09   95.49
#Mann= 3 , 0 , 0
       0    .055       0   42.87    .035       0   47.47    .055       0
Bank Sta=42.87,47.47
XS Rating Curve= 0 ,0
Exp/Cntr=0.3,0.1

Type RM Length L Ch R = 1 ,79.14   ,5.7,6.39,8.69
XS GIS Cut Line= 6
344172.5156860355422797.38391113344184.6442871095422820.23950195
344189.4959106455422830.80151367344192.6146850595422836.86169434
 344198.505676275422838.07373047344222.416687012 5422829.4163208
#Sta/Elev= 28
       0    97.1     .01    97.1   25.05   96.24   25.87   95.83    32.9   92.27
   34.18   91.47    37.5   90.71   37.59   90.69   38.88    90.5   39.24   90.38
   43.48   87.68   44.31   87.19   44.77    86.9   45.02   86.74   45.24   86.76
   46.21   86.73   46.81    86.8   47.05   86.79   47.47   86.88   47.98   86.97
   50.33   87.37   51.24   87.61   57.01   88.77   60.07   90.49   61.37   91.24
   66.36   94.17   72.64   94.49   75.76   94.63
#Mann= 3 , 0 , 0
       0    .055       0   44.77    .035       0   47.98    .055       0
Bank Sta=44.77,47.98
XS Rating Curve= 0 ,0
Exp/Cntr=0.3,0.1

Type RM Length L Ch R = 1 ,72.74   ,2.71,4.99,10
XS GIS Cut Line= 6
344171.8225097665422799.11547852344184.1245117195422820.93212891
344188.6295166025422839.97851563344193.3076782235422843.78771973
344216.6989135745422842.22930908344227.2681274415422834.95709229
#Sta/Elev= 19
       0   97.04   23.65   96.26   30.25    92.9   32.42   91.49   38.36    90.1
   45.04   88.05   47.79  86.196   48.14   85.96   51.41   86.04   52.44   86.18
   56.09   86.69   57.64   86.63   61.27   87.56   64.46   89.61   70.49   93.88
   71.28   93.99   75.63   94.03   84.82   94.49   86.94   94.73
#Mann= 3 , 0 , 0
       0    .055       0   47.79    .035       0   52.44    .055       0
Bank Sta=47.79,52.44
XS Rating Curve= 0 ,0
Exp/Cntr=0.3,0.1

Type RM Length L Ch R = 1 ,67.75   ,2.94,3.71,5.31
XS GIS Cut Line= 5
344170.9561157235422800.32751465344182.3919067385422821.62469482
344188.1096801765422845.86547852344201.4512939455422856.25427246
344215.1395263675422858.85168457
#Sta/Elev= 27
       0   96.98    3.31   96.96   22.52    96.3   24.17   95.47   28.09   93.47
   31.11   91.51   35.87    90.4   36.19   90.28    38.9   89.55   48.29   86.66
   49.08    86.4   49.29   86.34   50.28   85.67   50.92   85.24   55.32   85.35
   55.94   85.37   56.12   85.36   58.28   85.46   59.78   87.57   60.83   88.77
   62.39   90.67   62.61      91   65.25    92.8   65.99   92.96   66.38   93.03
   72.89    93.3   79.92   93.41
#Mann= 3 , 0 , 0
       0    .055       0   50.28    .035       0   55.32    .055       0
Bank Sta=50.28,55.32
XS Rating Curve= 0 ,0
Exp/Cntr=0.3,0.1

Type RM Length L Ch R = 1 ,64.04   ,3.68,3.35,4.35
XS GIS Cut Line= 5
344169.7432861335422800.50048828344180.4859008795422821.27832031
344182.5651245125422830.97467041344185.8572998055422847.59692383
344200.5848999025422866.29711914
#Sta/Elev= 27
       0   96.95    6.05    96.9   22.56   96.34   23.39   95.92   27.06   94.05
   30.93   91.53   33.31   90.97    34.4   90.72   34.92   90.53   39.51   89.28
   50.25   85.97   51.74   85.58   53.17    85.2   53.39   85.13   54.06    84.7
   56.42   84.67   56.83    84.7   57.07   84.72   59.16   85.17   62.57   89.71
   62.64   89.81   62.73   89.92   63.32   90.84   64.14   92.12    64.2   92.13
   66.17   92.54   74.06   92.49
#Mann= 3 , 0 , 0
       0    .055       0   53.39    .035       0   59.16    .055       0
Bank Sta=53.39,59.16
XS Rating Curve= 0 ,0
Exp/Cntr=0.3,0.1

Type RM Length L Ch R = 1 ,60.69   ,4.56,3.94,4.31
XS GIS Cut Line= 5
344164.1987304695422804.13671875344179.4462890635422833.39868164
 344182.738281255422847.25067139344187.9362792975422857.12011719
344197.6392822275422868.20172119
#Sta/Elev= 27
       0   96.71   18.01   96.56   20.34   96.48   21.09    96.1    28.4   91.58
   29.05   91.43   30.29   91.03      33   90.35   38.48   88.87   47.23   86.18
   50.88   85.13   52.04    84.8   53.43   84.34   55.58   84.69   55.79   84.72
   56.44   84.85   58.39   85.29   58.71   85.36   59.59   86.31   60.14   86.85
   61.16   88.51   63.18   91.86   64.13   91.99   64.96   92.34   65.02   92.35
   66.87   92.33   73.12   92.32
#Mann= 3 , 0 , 0
       0    .055       0   50.88    .035       0   55.58    .055       0
Bank Sta=50.88,55.58
XS Rating Curve= 0 ,0
Exp/Cntr=0.3,0.1

Type RM Length L Ch R = 1 ,56.76   ,7.72,5.83,4.41
XS GIS Cut Line= 4
344158.3076782235422827.16552734 344178.579895025422847.07751465
344186.7235107425422864.21929932344193.4810791025422870.10632324
#Sta/Elev= 23
       0   96.48    5.04    96.4    8.11   93.83   11.37   92.34   15.68   89.62
   18.36   88.67   21.86   87.95   28.42   86.38   31.19   85.57   33.47   84.81
   35.37   84.17   38.73   84.71   40.25   84.96   41.38   85.13   42.15   87.01
   43.35    87.9   44.82   90.58   44.99   90.62   46.16   91.45   47.39   91.98
   47.99   92.23   48.26   92.31   56.36    92.2
#Mann= 3 , 0 , 0
       0    .055       0   33.47    .035       0   38.73    .055       0
Bank Sta=33.47,38.73
XS Rating Curve= 0 ,0
Exp/Cntr=0.3,0.1

Type RM Length L Ch R = 1 ,50.93   ,7.48,7.07,7.18
XS GIS Cut Line= 3
344154.1492919925422830.97467041344182.045288086 5422862.4876709
344192.0949096685422870.62567139
#Sta/Elev= 27
       0   96.43    4.55   96.35    5.62   95.45    8.95   93.95    9.45   93.86
   12.53   91.66   14.82   90.06   19.75   87.21   20.66   86.81   21.68   86.49
   27.38   84.93   28.89   84.55   30.17  84.189   30.91   83.98   31.27   83.88
   31.63   83.94   36.01   84.58   38.61   84.95   40.23   88.54   41.68   90.29
   42.09   90.24   42.78   90.17   44.72   91.09   45.71    91.8    46.7   92.19
   47.04    92.3   55.02   92.19
#Mann= 3 , 0 , 0
       0    .055       0   30.17    .035       0   36.01    .055       0
Bank Sta=30.17,36.01
XS Rating Curve= 0 ,0
Exp/Cntr=0.3,0.1

Type RM Length L Ch R = 1 ,43.86   ,6.35,6.86,7.11
XS GIS Cut Line= 3
344148.4312744145422837.38128662344180.3126831055422869.93310547
344188.4562988285422875.99328613
#Sta/Elev= 21
       0   96.52    4.55   95.97   12.51   89.96   12.71   89.84   14.08   88.75
   14.25   88.65   14.38   88.55   26.94  83.804   27.48    83.6   27.99   83.54
   28.02   83.54   28.14   83.59   33.56   84.03   35.67    84.2   39.14   88.33
   41.47   89.96   45.36    92.2   45.56    92.2   47.15   92.23   50.35   92.17
   55.71    92.1
#Mann= 3 , 0 , 0
       0    .055       0   26.94    .035       0   33.56    .055       0
Bank Sta=26.94,33.56
XS Rating Curve= 0 ,0
Exp/Cntr=0.3,0.1

Type RM Length L Ch R = 1 ,37.00   ,27.23,24.86,22.79
XS GIS Cut Line= 3
344145.4793090825422841.12591553344173.7730712895422874.27587891
 344184.958923345422878.58673096
#Sta/Elev= 19
       0   96.14    4.25   95.62    8.93   92.07   10.99   90.63   13.32   90.19
   13.73   89.97   18.66   86.27    25.7   83.58   27.09   83.43   29.82   83.13
   30.72   83.51   32.12   83.62    33.8   83.75   35.14   85.35   43.58   91.17
   44.18   91.57   45.06   92.04   50.26   92.15   55.57   92.07
#Mann= 3 , 0 , 0
       0    .055       0   27.09    .035       0   32.12    .055       0
Bank Sta=27.09,32.12
XS Rating Curve= 0 ,0
Exp/Cntr=0.3,0.1

Type RM Length L Ch R = 1 ,12.14   ,4.7,12.15,6.96
XS GIS Cut Line= 6
344139.0648803715422843.84472656344136.9857177735422848.86608887
344142.5302734385422874.31890869344145.1292724615422880.89849854
344157.6044921885422887.30487061344184.6342773445422879.51330566
#Sta/Elev= 29
       0    96.1    5.43   95.84    5.48   95.84   13.26   92.56   14.37    91.9
   15.84   91.54   17.28   91.32   21.12   90.73   25.12   89.93   29.84   88.78
   31.48   87.72   31.88   87.46   34.77   85.25   38.56   82.95   39.11  82.606
   39.52   82.35    40.9   82.42   45.09   82.63   46.48   82.65   47.95   82.68
   50.31   84.26   52.58   85.06   57.87   87.62    58.5   87.85   63.47   89.97
   63.73   90.05   70.56   91.99   74.61    92.1   80.71   92.06
#Mann= 3 , 0 , 0
       0    .055       0   39.11    .035       0   45.09    .055       0
Bank Sta=39.11,45.09
XS Rating Curve= 0 ,0
Exp/Cntr=0.3,0.1

River Reach=BellsB          ,M002
Reach XY= 30
342253.7468872075421134.60931396342350.9110717775421129.54528809
342443.6716918955421244.12451172342442.2005004885421466.38751221
342499.714477539  5421578.284729342582.4801025395421661.34710693
342588.6450805665421717.04992676342637.0739135745421745.06988525
342593.8115234385421952.46270752342607.6630859385422009.07128906
342568.2431030275422041.64990234342629.994873047 5422104.3192749
 342599.371093755422241.19927979342679.5280761725422369.15911865
342764.2416992195422389.19268799342898.6043090825422369.78991699
342973.2835083015422459.28948975343043.7155151375422683.67950439
343121.2028808595422725.05749512343206.7385253915422666.71209717
343299.5507202155422773.61712646343475.9014892585422722.18811035
343520.2786865235422782.17248535343600.3688964845422818.95428467
343699.2672729495422816.61627197 343718.119079595422849.35510254
343842.1005249025422833.88592529343938.5328979495422872.97729492
343987.3618774415422852.26452637344144.2833251955422894.11730957

Type RM Length L Ch R = 1 ,5166.11 ,15.85,16.88,18.06
XS GIS Cut Line= 2
342277.9199218755421174.32928467342246.3927001955421094.99212646
#Sta/Elev= 21
       0  194.87    4.87  193.53    5.46  193.51   16.24  192.65    24.2  192.33
   30.49  193.13   33.24   192.5   35.69  191.76   36.61  191.67   44.35  191.12
   46.35  190.98   47.49  190.89   48.76 191.067   51.01  191.38   57.79  192.95
   61.01  193.34   61.28  193.35   67.04  193.71   80.92  194.96   81.94   195.1
   85.37  195.66
#Mann= 3 , 0 , 0
       0    .065       0   46.35     .04       0   48.76    .065       0
Bank Sta=46.35,48.76
XS Rating Curve= 0 ,0
Exp/Cntr=0.3,0.1

Type RM Length L Ch R = 1 ,5149.23 ,31.28,31.78,26.26
XS GIS Cut Line= 3
342284.6198730475421175.58990479342286.6940917975421159.00872803
 342266.990295415421094.41052246
#Sta/Elev= 21
       0  195.47    3.49  193.81    3.84   193.8   16.71   193.3   25.53  192.92
   29.75  192.59   30.83  192.56   32.16  192.51   37.45  191.29   43.45 190.867
   46.25  190.67   47.35  190.89   49.51  191.32   51.06  191.63   58.15  193.33
   58.71  193.48   63.94  193.76   64.25  193.76   64.35  193.77   65.97  193.87
   84.25  195.04
#Mann= 3 , 0 , 0
       0    .065       0   43.45     .04       0   47.35    .065       0
Bank Sta=43.45,47.35
XS Rating Curve= 0 ,0
Exp/Cntr=0.3,0.1

Type RM Length L Ch R = 1 ,5117.45 ,19.84,26.6,30.57
XS GIS Cut Line= 3
342310.9426879885421195.21392822342324.6160888675421164.53149414
342286.500915527  5421097.578125
#Sta/Elev= 22
       0  194.13   25.55  193.85   33.59   194.1   38.54  194.16   41.05  193.98
   50.37  192.64   55.56  192.13   57.66   191.8   62.74 190.128    63.1  190.01
   64.68 190.056   69.63   190.2   71.63  190.26   72.67  190.29   81.52  191.19
   85.37  192.19   88.35  192.79    88.8  192.82    89.2  192.89   90.21  192.41
   92.38  192.75  110.63  193.96
#Mann= 3 , 0 , 0
       0    .065       0   62.74     .04       0   64.68    .065       0
Bank Sta=62.74,64.68
XS Rating Curve= 0 ,0
Exp/Cntr=0.3,0.1

Type RM Length L Ch R = 1 ,5090.85 ,11.72,23.38,30.25
XS GIS Cut Line= 5
342312.2744750985421195.62567139342333.3610839845421161.42669678
342330.595703125 5421119.2824707 342333.706909185421078.17468262
342337.5092773445421065.39331055
#Sta/Elev= 27
       0   194.1   22.87  193.79   40.18  194.32   41.65  194.36   47.43  193.94
   53.42  193.07   56.52  191.95   68.58  190.24   69.99     190   71.67  189.72
   72.07   189.9   76.71  192.03   78.35  192.54   79.25  193.21   79.73  193.31
   80.68  193.35   82.41  193.39  108.53  193.95  112.89  194.13  118.19  195.39
  119.36  195.97  120.17  196.21  123.64  196.42  123.87  196.44  125.17   196.4
  133.58  197.27  136.97  197.94
#Mann= 3 , 0 , 0
       0    .065       0   69.99     .04       0   72.07    .065       0
#XS Ineff= 2 , 0
       0   41.65  194.36               0
Permanent Ineff=
       F       F
Bank Sta=69.99,72.07
XS Rating Curve= 0 ,0
Exp/Cntr=0.3,0.1

Type RM Length L Ch R = 1 ,5067.47 ,48.56,49.69,45.53
XS GIS Cut Line= 4
342313.2647094735421195.98748779342339.321716309 5421161.1796875
342343.9644775395421135.16009521342390.2396850595421118.28967285
#Sta/Elev= 28
       0  194.08   21.43  193.76   43.48  194.43   44.88  194.47   53.25  193.91
   54.99  193.68   55.73  193.41   57.98  193.15   59.14  192.97      63  192.04
   69.91  190.81   71.59  190.71   74.24  189.32   77.36   189.3   78.38  189.28
   79.36   189.3   81.97  189.31   83.39  190.15   84.24   190.4   84.95  190.83
   87.31  191.88   89.04  192.69   95.49  192.94   96.14  192.88   99.25  192.84
  105.49  192.56  109.43  193.46  119.17  194.07
#Mann= 3 , 0 , 0
       0    .065       0   77.36     .04       0   79.36    .065       0
#XS Ineff= 2 , 0
       0   44.88  194.47               0
Permanent Ineff=
       F       F
Bank Sta=77.36,79.36
XS Rating Curve= 0 ,0
Exp/Cntr=0.3,0.1

Type RM Length L Ch R = 1 ,5017.78 ,49.08,50.21,50
XS GIS Cut Line= 3
 342317.392517095421198.30810547342365.3787231455421178.71252441
342418.3422851565421133.77050781
#Sta/Elev= 24
       0  194.11   18.61  194.11   39.21  194.11   51.83  194.09   63.38  194.18
   63.57  194.08   64.28  193.73    71.6  189.27   74.56  188.62   75.65  188.42
   76.84  188.22   77.65   188.3   83.16  188.89   84.81  189.71   86.95  190.68
   87.54  191.09   87.92  191.33   89.35   192.3   92.31  193.42   95.07  194.66
   97.02  194.78   106.3  195.04  111.18  195.38  121.29  195.93
#Mann= 3 , 0 , 0
       0    .065       0   75.65     .04       0   77.65    .065       0
#XS Ineff= 2 , 0
       0   63.38  194.18               0
Permanent Ineff=
       F       F
Bank Sta=75.65,77.65
XS Rating Curve= 0 ,0
Exp/Cntr=0.3,0.1

Type RM Length L Ch R = 1 ,4967.57 ,45.92,50.1,48.87
XS GIS Cut Line= 6
342356.3491210945421232.34228516342385.2438964845421220.99768066
342427.9514770515421189.73413086342426.5952758795421173.13287354
 342416.976684575421160.14831543342421.3626708985421134.88031006
#Sta/Elev= 28
       0  194.49   24.59  193.83    25.1  193.66   27.15  193.71   31.04  193.56
   40.92  193.16   47.29  189.87   52.49   187.2   53.57  186.65   54.49  186.78
   55.45  186.91   58.38  187.51   64.24  191.22   65.84  191.81   66.05   191.9
   72.02  192.65   83.97  192.17   87.42  192.03   91.08   192.8  100.63  193.39
  108.69  193.98  113.27  194.54  116.79  194.68  129.77  195.28   132.6   195.5
  137.39  195.53   141.9  195.98  142.43     196
#Mann= 3 , 0 , 0
       0    .065       0   52.49     .04       0   54.49    .065       0
Bank Sta=52.49,54.49
XS Rating Curve= 0 ,0
Exp/Cntr=0.3,0.1

Type RM Length L Ch R = 1 ,4917.46 ,19.17,44.16,54.69
XS GIS Cut Line= 6
342357.8818969735421262.62231445 342432.634704595421247.08508301
342461.317871094 5421216.9163208342469.8649291995421203.72247314
342491.2780761725421192.89349365342526.8798828135421141.00531006
#Sta/Elev= 23
       0  194.19   40.11  193.67   49.66  191.92   55.26  188.11   56.48  187.75
   67.37  186.39   76.23  188.14   76.67  188.12   77.24  187.96   82.26  185.81
   83.82  185.79   85.67  185.87   91.56  185.89   92.94  186.53   99.38  190.01
  148.09  189.96  151.23  190.19  162.06  190.26  169.52  190.43  193.67  192.13
  210.51  194.03  213.95  194.31  220.62   194.6
#Mann= 3 , 0 , 0
       0    .065       0   82.26     .04       0   85.67    .065       0
Bank Sta=82.26,85.67
XS Rating Curve= 0 ,0
Exp/Cntr=0.3,0.1

Type RM Length L Ch R = 1 ,4873.31 ,21.46,19.89,10.45
XS GIS Cut Line= 4
342358.6434936525421270.36907959342438.6124877935421267.15551758
342445.2736816415421278.15710449342491.5441284185421265.21850586
#Sta/Elev= 30
       0  194.11    35.5  193.61   37.89  193.54   43.94  193.08   47.42  192.44
   55.33  187.31   55.68  187.19   66.45  187.35   73.94  186.69   76.96  186.27
   80.03  186.81   81.22  186.78   85.82  184.88   86.08  184.76   86.44  184.76
   87.82   185.2   89.97  185.87   94.68  187.08  101.43  187.22   105.2  188.17
  106.36  188.63  107.34  188.82  114.35  191.27  117.64  191.51  120.79  190.67
   123.7  190.95  126.56  190.92  132.13  193.27  134.49  193.35  140.94     194
#Mann= 3 , 0 , 0
       0    .065       0   85.82     .04       0   87.82    .065       0
Bank Sta=85.82,87.82
XS Rating Curve= 0 ,0
Exp/Cntr=0.3,0.1

Type RM Length L Ch R = 1 ,4853.42 ,50.5,50.5,50.5
XS GIS Cut Line= 4
342365.0905151375421337.63391113342412.5452880865421300.91088867
342419.1926879885421287.99310303342493.4204711915421266.96832275
#Sta/Elev= 26
       0     194   33.33     191   60.19     190   63.84     189   66.81     188
   69.53     187   73.96     186   78.15     186   80.75     185   82.02  184.06
   82.89  183.55   83.22  183.62   83.62  183.67   84.34  183.76   84.64  183.95
   90.18   184.6   91.54  184.71   96.24     186  100.78     187  106.81     188
  111.06     189   116.3     190  118.77     191  122.39     192  140.17     194
  151.68     195
#Mann= 3 , 0 , 0
       0    .065       0   82.02     .04       0   84.64    .065       0
#XS Ineff= 2 , 0
       0   82.02  193.62   84.42       0  193.62
Permanent Ineff=
       F       F
Bank Sta=82.02,84.64
XS Rating Curve= 0 ,0
Exp/Cntr=0.5,0.3

Type RM Length L Ch R = 2 ,4850    ,,,
BEGIN DESCRIPTION:
Ring Road (Structure #2129)
END DESCRIPTION:
Bridge Culvert--1,0,-1,-1, 0
Deck Dist Width WeirC Skew NumUp NumDn MinLoCord MaxHiCord MaxSubmerge Is_Ogee
17.25,12.2,1.67,0, 13, 13, 193.62, , 0.98, 0, 0.64,0.63,,
       0   18.35   68.32   74.04   77.93   81.43   84.94   88.48   92.35   95.81
  100.27  117.15  151.68
     194     194  193.66  193.62  193.64  193.64  193.66  193.74   193.8  193.87
  193.95     194     195
                                                                                
                        
       0     6.5   44.14   47.78   51.11    54.7   58.32   61.86   65.29   68.91
   73.04   98.35  139.95
     194     194  193.02  192.99  192.96  192.98  192.97  193.01  193.08  193.14
  193.06     194     195
                                                                                
                        
BR Coef=-1 , 0 , 0 ,, 0 ,,,0.8,-1,,0,
WSPro=,,,, 1 ,,,, 0 ,,,, 0 ,,,,-1 ,-1 ,-1 , 0 , 0 , 0 , 0 , 0
Culvert=1,2.4,,45.5,0.03,0.9,1,1,1,183.62,83.22,182.06,62.72,Culvert #1  , 0 ,2.3
Culvert Bottom n=0.03
BC Design=,, 0 ,, 0 ,,,,,,
BC Use User HTab Curves=0
BC User HTab FreeFlow(D)= 0

Type RM Length L Ch R = 1 ,4805.77 ,17.89,20,21.25
XS GIS Cut Line= 6
      342378.992     5421357.995      342408.049      5421341.11
      342423.395      5421336.35      342441.668     5421333.993
      342441.668     5421333.993      342503.085     5421296.461
#Sta/Elev= 27
       0     194    4.62     193   15.63     192    34.9     190    41.9     188
   45.96     186    48.8     185   54.42     184   56.37  183.86   60.21  182.58
   60.84  181.97   61.59  181.72   62.72  181.53   64.55  182.13   65.21     183
   65.83  183.17    67.2  183.89   68.87     185   70.59  185.61   73.05     186
   81.24     187   90.22     188   96.57     189  110.06     190  134.12     191
   139.5     192  139.95     195
#Mann= 3 , 0 , 0
       0    .057       0   60.84     .04       0   64.55    .057       0
#XS Ineff= 2 , 0
       0   61.52   189.5   63.92       0   189.5
Permanent Ineff=
       F       F
Bank Sta=60.84,64.55
XS Rating Curve= 0 ,0
Exp/Cntr=0.5,0.3

Type RM Length L Ch R = 1 ,4785.76 ,29.07,29.11,29.57
XS GIS Cut Line= 4
342381.8477172855421362.48071289342405.0465087895421351.04650879
 342451.236511235421353.20410156342487.4505004885421330.52331543
#Sta/Elev= 23
       0  191.79   11.47   190.1   11.65  190.08   11.78  190.07   11.92  190.05
   13.91  189.77   25.86  188.34   27.17  188.12    53.6  181.71    54.2 181.581
   54.58   181.5    55.1  181.52    57.1   181.6   57.25   181.6   58.13  181.96
   61.53  184.66   62.79   185.1   62.85  185.12   66.84  185.01   70.98  185.32
    72.1  185.38   89.47  186.85  114.83  188.92
#Mann= 3 , 0 , 0
       0    .057       0    54.2     .04       0    57.1    .057       0
Bank Sta=54.2,57.1
XS Rating Curve= 0 ,0
Exp/Cntr=0.3,0.1

Type RM Length L Ch R = 1 ,4756.65 ,30.95,29.11,26.42
XS GIS Cut Line= 3
342393.0432739265421378.32452393342446.4367065435421382.54150391
342470.5885009775421367.50811768
#Sta/Elev= 20
       0  188.53    9.27  187.54   18.62  185.87   20.92  185.56   28.55  181.82
   30.15  181.09   33.92  180.71   37.43 180.352   38.72  180.22   38.83  180.21
      39  180.25   39.68   180.4   40.13   180.5      41  180.64   53.56   182.7
   64.04  184.27   65.91  184.34   68.17  184.59    72.8  184.92   82.01  185.68
#Mann= 3 , 0 , 0
       0    .057       0   37.43     .04       0   39.68    .057       0
Bank Sta=37.43,39.68
XS Rating Curve= 0 ,0
Exp/Cntr=0.3,0.1

Type RM Length L Ch R = 1 ,4727.54 ,19.26,20,19.72
XS GIS Cut Line= 4
342396.6063232425421408.54730225342417.0162963875421413.36407471
342443.3679199225421407.66790771342470.1505126955421385.22271729
#Sta/Elev= 22
       0  186.73    4.63  186.04    6.12  185.87    6.93  185.74   15.09  184.56
   20.97  183.26   24.07  182.65    26.6  181.37   30.23  179.76   32.67  179.74
   34.33  179.65   36.61  179.53   42.07 179.225   44.84  179.07   45.24 179.254
   47.93  180.49   49.08  181.23   53.41  182.09   54.95  182.14    61.7  182.47
   75.76  184.04   82.88  184.57
#Mann= 3 , 0 , 0
       0    .057       0   42.07    .037       0   45.24    .057       0
Bank Sta=42.07,45.24
XS Rating Curve= 0 ,0
Exp/Cntr=0.3,0.1

Type RM Length L Ch R = 1 ,4707.54 ,5.01,5.31,4.99
XS GIS Cut Line= 3
342405.9539184575421428.78527832342427.0795288095421431.20550537
342478.2404785165421415.30487061
#Sta/Elev= 25
       0  184.77      .8  184.65    3.41  184.08   11.15  183.67   15.84  183.34
   16.68  183.26   16.74  183.25   21.26  180.85   21.27  180.85   21.89  180.52
   23.25  179.93   30.32  178.96   33.06  178.28   33.98  178.05   37.37  178.05
    38.6  178.03      40  178.01   42.46 178.064    49.2  178.21    52.4  179.92
   65.34  182.16   67.64  182.47   69.94  182.91   71.52  183.07   74.84  183.28
#Mann= 3 , 0 , 0
       0    .057       0   37.37    .037       0   42.46    .057       0
Bank Sta=37.37,42.46
XS Rating Curve= 0 ,0
Exp/Cntr=0.3,0.1

Type RM Length L Ch R = 1 ,4702.24 ,16.74,19.76,23.42
XS GIS Cut Line= 3
342405.385681152 5421433.7454834342427.5565185555421436.28552246
342479.7224731455421420.07269287
#Sta/Elev= 26
       0  184.64     .14  184.64    6.11  184.07   17.04  183.14   17.44   183.1
   18.41  182.89   22.32  180.69    23.2  180.19   23.51     180   25.32  179.87
   31.43  179.52   32.12  179.47   32.25  179.47   32.66  179.41   33.13  179.29
   36.37  177.95   36.94  177.71   40.39  177.97   41.34  177.99   52.12  178.24
   54.39  179.44   69.79  182.11   72.26  182.82   74.72  182.94   75.35  182.95
   76.94  183.01
#Mann= 3 , 0 , 0
       0    .057       0   36.37    .037       0   40.39    .057       0
Bank Sta=36.37,40.39
XS Rating Curve= 0 ,0
Exp/Cntr=0.3,0.1

Type RM Length L Ch R = 1 ,4682.48 ,24.78,23.69,17.54
XS GIS Cut Line= 3
342384.6652832035421449.13708496342462.1015014655421451.67608643
342490.3955078135421431.71368408
#Sta/Elev= 21
       0  184.23    6.08  183.17    7.27  183.08    27.1  183.85   40.25  182.68
   40.66  182.59   42.69  181.43   45.75  179.52   49.09  179.24   49.65  179.13
   55.24 176.766   55.42  176.68   59.29  176.91   67.95  177.33   77.48   178.4
   83.28  178.87   88.85  180.58   90.14  180.79   92.25   181.5   97.37  181.89
  112.11  182.74
#Mann= 3 , 0 , 0
       0    .057       0   55.24    .037       0   59.29    .057       0
Bank Sta=55.24,59.29
XS Rating Curve= 0 ,0
Exp/Cntr=0.3,0.1

Type RM Length L Ch R = 1 ,4658.79 ,20.47,25.37,24.27
XS GIS Cut Line= 4
342413.6375122075421476.55328369342443.7119140635421474.82592773
 342454.427917485421468.95349121342486.5764770515421446.49951172
#Sta/Elev= 21
       0  183.73   14.57     183   17.96  181.58   23.03  177.93   24.07  177.84
   30.12  176.43   31.78  175.78   32.09  175.59   33.83  175.55   34.06  175.55
    34.4  175.73   37.22  177.27   38.05  177.54   39.65  177.77   46.28  178.19
   50.19  178.31   57.87  178.75   65.04  179.53    65.9  179.53   69.41  180.72
   81.56  181.64
#Mann= 3 , 0 , 0
       0    .057       0   31.78    .037       0    34.4    .057       0
Bank Sta=31.78,34.4
XS Rating Curve= 0 ,0
Exp/Cntr=0.3,0.1

Type RM Length L Ch R = 1 ,4633.41 ,27.81,23.8,18.32
XS GIS Cut Line= 4
342416.7960815435421491.53570557342437.1434936525421493.58789063
342478.5769042975421484.43591309342504.669311523 5421459.3939209
#Sta/Elev= 25
       0  183.21   13.96  182.53   17.01  180.89   20.45  180.15   24.58  178.73
   28.12  177.31   29.03  177.03   29.55  176.87   36.76  176.05   38.89  175.38
   47.43  174.88   49.43  174.77   50.68 174.697   52.17  174.61   52.47  174.56
   52.79  174.66   53.59  174.98   58.46  177.06    59.2  177.48   62.88  177.18
   63.67  177.12   68.66  177.81   74.47   179.5   84.38  180.18   99.05  181.43
#Mann= 3 , 0 , 0
       0    .057       0   50.68    .037       0   52.79    .057       0
Bank Sta=50.68,52.79
XS Rating Curve= 0 ,0
Exp/Cntr=0.3,0.1

Type RM Length L Ch R = 1 ,4609.61 ,24.92,25.62,25.97
XS GIS Cut Line= 5
342429.1931152345421518.69750977342463.0698852545421519.04290771
342476.8972778325421500.38891602342476.5516967775421488.98931885
342508.7000732425421460.66271973
#Sta/Elev= 29
       0  181.93    3.62  181.76    7.25  180.64   19.36  180.42   30.09  179.73
   33.88  179.41   38.21  179.29   39.09  179.12   44.66  174.94   45.98   173.9
   46.55   173.8   48.75  173.66   50.58  173.55   50.77  173.54   50.82  173.55
   51.53 173.666    54.5  174.15    57.1  174.78   64.98  176.92   65.12  176.95
   66.47  177.06    68.5  177.22   70.92  177.24    71.3  177.25   74.13  177.04
   77.52  177.49   84.07   179.4   95.67  180.19  111.35  181.51
#Mann= 3 , 0 , 0
       0    .057       0   48.75    .037       0   51.53    .057       0
Bank Sta=48.75,51.53
XS Rating Curve= 0 ,0
Exp/Cntr=0.3,0.1

Type RM Length L Ch R = 1 ,4583.99 ,44.18,49.27,61.24
XS GIS Cut Line= 3
342431.0048828135421538.47949219342482.4049072275421532.46948242
342524.3275146485421484.73327637
#Sta/Elev= 19
       0  181.46    2.43  181.36    2.96  181.19    6.88  181.03   45.97  178.36
   48.92   177.6   58.76   176.5   62.54   173.3   63.31  172.82      64  172.84
   65.52  173.29   68.29  174.14   72.46  174.97   83.74  175.17   90.83  177.19
   93.45  178.29  109.24   179.8  111.57  180.09  115.28  180.36
#Mann= 3 , 0 , 0
       0    .057       0   62.54    .037       0   65.52    .057       0
Bank Sta=62.54,65.52
XS Rating Curve= 0 ,0
Exp/Cntr=0.3,0.1

Type RM Length L Ch R = 1 ,4534.72 ,52.34,49.2,34.25
XS GIS Cut Line= 6
342436.604125977 5421544.3560791  342456.17968755421542.00231934
342507.2526855475421565.09869385342533.8956909185421539.60070801
342533.8956909185421523.66491699342551.0834960945421500.07147217
#Sta/Elev= 25
       0  180.92   19.72  179.74   47.53  177.21   53.12  175.92   58.77  171.71
   61.31  170.19   61.87  170.05   62.56  170.18   69.48  171.57   75.77  171.49
   84.93  171.86   94.04  174.51    96.1  174.64   99.35  175.81  100.58  175.95
  108.94  176.42  112.74  176.16  114.11  177.01  123.21  177.01  124.19  177.12
  129.59   177.3   131.7   177.3  135.88  177.61  143.88  179.07  158.78  179.81
#Mann= 3 , 0 , 0
       0    .057       0   61.31    .037       0   62.56    .057       0
Bank Sta=61.31,62.56
XS Rating Curve= 0 ,0
Exp/Cntr=0.3,0.1

Type RM Length L Ch R = 1 ,4485.52 ,46.5,49.24,52.08
XS GIS Cut Line= 4
342476.4520874025421609.90167236342512.644287109 5421605.4152832
342558.8079223635421563.58587646 342569.720886235421526.56231689
#Sta/Elev= 21
       0  176.02    4.81  176.04   13.03  174.17      16  173.93   41.51  170.86
   45.37  169.57   47.78 168.396   48.08  168.25   50.46  168.32    61.7  168.67
   76.06  169.53   77.43  169.73   80.16  170.75   89.65  174.01   92.21  174.45
   95.66  174.69  106.19  175.11  125.01  176.84  129.12   176.9  131.74  177.36
  137.36  177.79
#Mann= 3 , 0 , 0
       0    .057       0   47.78    .037       0   50.46    .057       0
Bank Sta=47.78,50.46
XS Rating Curve= 0 ,0
Exp/Cntr=0.3,0.1

Type RM Length L Ch R = 1 ,4436.28 ,49.6,49.24,49.91
XS GIS Cut Line= 2
342514.9763183595421651.73468018342609.2982788095421603.30792236
#Sta/Elev= 18
       0  173.17    2.59  172.57    4.35  171.46     7.3  170.81   23.01   169.7
   30.77  168.23   33.48  167.98   39.63  166.85   47.26  166.03   49.18   165.9
   49.54 166.001   53.22  167.06   66.62  167.22   79.33  169.01   91.03  169.57
   93.72  170.25  105.12  172.57  106.03  172.61
#Mann= 3 , 0 , 0
       0    .057       0   47.26    .037       0   49.54    .057       0
Bank Sta=47.26,49.54
XS Rating Curve= 0 ,0
Exp/Cntr=0.3,0.1

Type RM Length L Ch R = 1 ,4387.04 ,46.3,49.24,50.07
XS GIS Cut Line= 5
342529.6284790045421685.46728516342563.0474853525421672.84527588
342570.367919922 5421677.3192749342608.3071289065421658.34008789
342632.8118896485421651.14147949
#Sta/Elev= 26
       0  174.04    3.06  173.53   12.01  172.33   15.57  171.26      22  168.14
   22.75  168.03    23.9  168.03   26.97  169.18   33.04  171.15    38.9  170.96
   47.31   170.3   50.14   168.7   55.58  166.81   59.96   164.4   61.19  164.21
   62.09  164.11   63.19  164.28   66.23  164.73    79.2  166.28   90.75  166.39
   92.49  166.92    93.2  166.93   99.79   168.1  104.38  169.17  108.41  171.72
  112.26  173.91
#Mann= 3 , 0 , 0
       0    .057       0   61.19    .037       0   63.19    .057       0
Bank Sta=61.19,63.19
XS Rating Curve= 0 ,0
Exp/Cntr=0.3,0.1

Type RM Length L Ch R = 1 ,4337.80 ,50.62,49.24,33.92
XS GIS Cut Line= 3
342552.150695801 5421724.3861084342620.3140869145421706.85028076
342649.2227172855421690.75970459
#Sta/Elev= 26
       0  172.48    1.81  172.33     2.3  172.07    4.45  171.21     7.9   169.6
    9.21  169.27   20.56  167.22   26.56  165.92   27.28  165.68      29  165.58
   36.17  162.89   36.78  162.65   38.17  162.79   45.13  163.47   50.19  163.71
   57.67  164.26   64.65  164.24   70.38  163.45   72.09  163.29   73.24  163.36
   78.76  166.02   79.74  166.34   93.36  168.56   93.97  168.81   98.79  171.53
  103.47  174.57
#Mann= 3 , 0 , 0
       0    .057       0   36.17    .037       0   38.17    .057       0
Bank Sta=36.17,38.17
XS Rating Curve= 0 ,0
Exp/Cntr=0.3,0.1
