HEC-RAS study Corner_Brook2.prj: Corner_Brook2

--- Corner_Brook2.g02 (geometry) --- (continued)

Type RM Length L Ch R = 1 ,1848.27 ,12.45,13.99,15.17
XS GIS Cut Line= 3
343896.088500977 5422883.3649292343932.2098999025422838.39147949
343929.8264770515422826.35388184
#Sta/Elev= 26
       0  108.11    7.65  108.08   10.94  107.87   11.97   107.8   14.48  107.19
   25.17   99.99    35.5    92.8   35.82   92.43   37.95   92.51    38.5   92.45
    41.5   91.91   42.22   92.03   42.78  92.487   47.16   96.06   50.51   98.19
   51.76   99.15   53.45  100.46   56.58  100.74   57.57  100.77   57.68  100.78
   57.87  100.79   60.69  101.05   65.85   104.5    68.3  106.05   69.09   106.5
   69.95  106.51
#Mann= 3 , 0 , 0
       0     .06       0    38.5     .04       0   42.78     .05       0
Bank Sta=38.5,42.78
XS Rating Curve= 0 ,0
Exp/Cntr=0.3,0.1

Type RM Length L Ch R = 1 ,1834.27 ,15.6,12.92,10.12
XS GIS Cut Line= 4
343910.1044921885422880.51928711343924.2083129885422866.56329346
343938.5886840825422857.58172607343933.0576782235422839.61871338
#Sta/Elev= 24
       0  106.27    2.47  105.62    6.96  102.49    19.4   93.69   19.84   93.48
   22.57   92.19   23.56   91.67   24.52   91.16   26.57   90.88   27.65   91.72
   34.63   97.31   35.27   97.83   35.54   98.02    36.8   98.23   36.94   98.26
   37.15   98.23   37.65   98.08   37.99   98.12   39.13    98.6    47.9   99.51
   50.54  100.49   50.62   100.5   51.59   100.6   55.59  100.77
#Mann= 3 , 0 , 0
       0     .06       0   23.56     .04       0   27.65     .05       0
Bank Sta=23.56,27.65
XS Rating Curve= 0 ,0
Exp/Cntr=0.3,0.1

Type RM Length L Ch R = 1 ,1821.35 ,17.76,13.93,9.68
XS GIS Cut Line= 5
 343926.697082525422893.36987305343934.9935302735422878.44671631
343940.5244750985422865.87249756343939.9713134775422860.20709229
343932.9194946295422838.65148926
#Sta/Elev= 30
       0  105.32     2.5  104.28    4.01  103.35    9.14   98.81   13.08   96.22
   15.87   93.87   17.07   93.17   18.17   92.56   20.82   91.15   22.07   91.14
   24.14    90.9   25.07   91.13   26.91   91.15   28.97   92.75   30.81   94.14
   32.26   95.32   33.93   96.33   35.74   97.34    36.5   97.56   38.73   98.16
   39.41   98.29   39.72   98.24   40.48   98.02   40.97   98.08   42.61   98.78
   50.48   99.56   52.95  100.47   54.03  100.61   54.14  100.62   59.18  100.82
#Mann= 3 , 0 , 0
       0     .06       0   22.07     .04       0   25.07     .05       0
Bank Sta=22.07,25.07
XS Rating Curve= 0 ,0
Exp/Cntr=0.3,0.1

Type RM Length L Ch R = 1 ,1807.43 ,6.99,6.66,6.33
XS GIS Cut Line= 4
343963.0629272465422890.60632324 343943.566528325422858.41088867
 343938.173889165422854.81829834343933.4724731455422838.78967285
#Sta/Elev= 28
       0   99.39    5.79   99.31    7.82   99.06   18.11   91.55    19.4   90.67
    19.6   90.53   21.59   90.32   23.95   90.07   24.67   89.83   25.15   90.38
   30.13   93.26   33.28   96.23   34.71   97.11   37.64   98.07   38.95   98.42
   39.27   98.46   39.39   98.47   40.66   98.29   42.45    97.9   43.12   98.02
   44.12   98.61    44.5   98.77   52.37    99.6   54.64  100.46   55.74   100.6
   56.21  100.61   56.64  100.66   60.82  100.85
#Mann= 3 , 0 , 0
       0     .06       0   21.59     .04       0   25.15     .05       0
Bank Sta=21.59,25.15
XS Rating Curve= 0 ,0
Exp/Cntr=0.3,0.1

Type RM Length L Ch R = 1 ,1800.77 ,20.94,22.78,23.41
XS GIS Cut Line= 2
343975.0184936525422892.67388916343935.345092773 5422837.5770874
#Sta/Elev= 25
       0   98.94    7.72   98.92      15   98.84   15.35    98.8   17.32   97.38
   20.73   95.07   26.19   91.35   26.87   90.88   28.67   90.62   30.17   90.39
   31.99  90.111   33.17   89.93   34.05   89.59   34.41    89.9   34.68  90.151
   38.88   94.06   42.23   96.61   48.48   97.06   51.82   97.09   52.73   97.23
   54.85   98.36   59.48  100.28   64.04  100.49   67.43  100.95   67.89  100.96
#Mann= 3 , 0 , 0
       0     .06       0   31.99     .04       0   34.68     .05       0
Bank Sta=31.99,34.68
XS Rating Curve= 0 ,0
Exp/Cntr=0.3,0.1

Type RM Length L Ch R = 1 ,1777.98 ,21.46,24.72,28.06
XS GIS Cut Line= 4
343980.1383056645422888.39147949343976.5432739265422857.16333008
343969.353088379 5422842.2401123343975.1605224615422812.39367676
#Sta/Elev= 21
       0   98.63   14.33   98.09   19.42   94.75   24.65   91.07   25.12   90.87
   29.94   89.43   31.43   89.25   32.26   89.17   34.42   88.77   35.43    89.4
    38.9   90.72   45.79   95.17      48   96.76   49.54   97.86   54.51   98.88
   54.85   99.01   55.63    99.2   61.03   99.98   61.85  100.13   77.47  102.82
   78.41  103.36
#Mann= 3 , 0 , 0
       0     .06       0   32.26     .04       0   35.43     .05       0
Bank Sta=32.26,35.43
XS Rating Curve= 0 ,0
Exp/Cntr=0.3,0.1

Type RM Length L Ch R = 1 ,1753.27 ,23.46,23.53,23.82
XS GIS Cut Line= 2
 343986.71307373 5422892.0324707344012.6475219735422816.35290527
#Sta/Elev= 22
       0   98.92   18.68   98.32   22.14   96.31   28.45   92.83   29.25   92.29
   32.77   90.77    38.5    88.7   39.25   88.22    41.5   89.07   42.91   89.47
   47.67   93.49   51.89   96.16    56.3   97.04   57.21      97   59.09   97.58
   62.73   98.53   65.88    99.8   67.81  100.49   71.29  102.33   71.32  102.34
   72.02  102.35      80  102.58
#Mann= 3 , 0 , 0
       0     .06       0    38.5     .04       0    41.5     .05       0
Bank Sta=38.5,41.5
XS Rating Curve= 0 ,0
Exp/Cntr=0.3,0.1

Type RM Length L Ch R = 1 ,1729.73 ,23.22,23.97,25.7
XS GIS Cut Line= 4
344003.0916748055422887.14788818344015.6744995125422879.13348389
344034.7561035165422826.34967041344033.2351074225422814.88092041
#Sta/Elev= 22
       0   98.35    3.45   98.22   13.56   97.57   14.92   97.45   15.28   97.44
    18.6   96.52   29.29   89.02   29.47   88.91   31.83   88.69   33.89  88.492
   35.21   88.17   36.78  88.572   39.18   88.88   39.19   88.89   47.64   93.81
   53.88   97.73   57.23   98.86   62.66  101.12   63.76  101.39   71.05  101.51
    82.3  101.93   82.61  101.94
#Mann= 3 , 0 , 0
       0     .06       0   33.89     .04       0   36.78     .05       0
Bank Sta=33.89,36.78
XS Rating Curve= 0 ,0
Exp/Cntr=0.3,0.1

Type RM Length L Ch R = 1 ,1705.77 ,17.93,16.86,16.52
Node Photo=..\..\..\..\Corner Brook\Windshield Survey\CB photos\P1000705.JPG
XS GIS Cut Line= 5
      344012.139     5422902.717      344019.302     5422901.315
       344026.26     5422902.924      344029.788     5422896.702
      344064.067     5422832.421
#Sta/Elev= 28
       0      98     8.8      97   14.44   96.22   21.54   95.94    30.3   95.92
   30.41   95.91   32.85   95.66   33.78   95.64   34.05    95.5   39.56   92.22
   41.37    91.3   49.73   88.13   52.91   87.96   55.84    87.6    56.9  87.962
   62.86   88.87    63.9   89.02   64.48   89.24   64.86   89.36   65.86   89.75
    67.7   90.62    69.6   91.65   70.69   92.44   76.82   95.21   83.98   99.16
    85.9   99.87   86.12   99.88   94.44   99.85
#Mann= 3 , 0 , 0
       0     .06       0   52.91    .035       0    56.9    .055       0
Bank Sta=52.91,56.9
XS Rating Curve= 0 ,0
Exp/Cntr=0.3,0.1

Type RM Length L Ch R = 1 ,1688.91 ,64.88,64.59,65.49
XS GIS Cut Line= 5
      344005.862     5422920.796      344017.456     5422919.468
      344045.474     5422913.779      344048.045     5422907.328
       344072.87     5422838.617
#Sta/Elev= 27
       0      98   11.43      97   40.26      96   57.82      96   60.54      95
   62.12      94   63.41      93   65.14      92   66.69      91   70.08      90
   74.11   89.16   75.38      88   76.46   87.38   76.99   86.72   78.53   86.72
   79.32   87.09   80.66   86.92   81.21  87.996    81.8   89.15   84.75   89.15
   88.39      91   92.98      94   95.38      95  101.56      97  110.05      98
  113.44      99  120.26      99
#Mann= 3 , 0 , 0
       0     .06       0   75.38    .035       0   81.21    .055       0
#XS Ineff= 2 , 0
       0   76.73   95.43   78.53       0   95.43
Permanent Ineff=
       F       F
Bank Sta=75.38,81.21
XS Rating Curve= 0 ,0
Exp/Cntr=0.5,0.3

Type RM Length L Ch R = 2 ,1650    ,,,
BEGIN DESCRIPTION:
Bliss Street (Structure #2120)
END DESCRIPTION:
Bridge Culvert--1,0,-1,-1, 0
Deck Dist Width WeirC Skew NumUp NumDn MinLoCord MaxHiCord MaxSubmerge Is_Ogee
21.2,15.5,1.67,0, 11, 13, 95.43, , 0.98, 0, 0.7,0.53,,
   40.26   52.35   56.26   60.77   66.61   74.88   81.52   88.61   97.05  113.06
  120.26
   95.43   95.43   95.44   95.53   95.63   95.86    96.1   96.39   96.86      98
   97.38
                                                                                
        
       0   10.32   13.62   17.53   22.04   28.85   36.98   44.83   51.73   59.58
   67.12    75.2      80
      95      95   95.43   95.44   95.53   94.97   95.53   96.06   96.49   96.95
   97.28   97.38   97.38
                                                                                
                        
BR Coef=-1 , 0 , 0 ,, 0 ,,,0.8,-1,,0,
WSPro=,,,, 1 ,,,, 0 ,,,, 0 ,,,,-1 ,-1 ,-1 , 0 , 0 , 0 , 0 , 0
Culvert=1,1.8,,56,0.03,0.5,1,2,1,86.72,77.63,84.33,38.91,Culvert #1  , 0 ,4.4
Culvert Bottom n=0.03
BC Design=,, 0 ,, 0 ,,,,,,
BC Use User HTab Curves=0
BC User HTab FreeFlow(D)= 0

Type RM Length L Ch R = 1 ,1624.32 ,17.6,18.73,19.48
Node Photo=..\..\..\..\Corner Brook\Windshield Survey\CB photos\P1000701.JPG
XS GIS Cut Line= 2
344108.9406738285422918.89208984344136.3378906255422843.72967529
#Sta/Elev= 28
       0   93.51   10.08   93.51   23.42      93   24.64      92      26      91
   26.89      90   28.23      89   29.56      88   30.81      87   31.84      86
   33.38      85   34.32      84   38.91   83.97   46.21      84   47.63      85
   48.76      86   49.86      87   51.64      88   53.79      89   58.39      90
   59.97      91   63.23      92   65.08      93   67.45      94   69.57      95
   71.74      96   76.49   96.16      80   96.23
#Mann= 3 , 0 , 0
       0     .06       0   33.38    .035       0   47.63    .055       0
#XS Ineff= 2 , 0
       0   38.01   90.55   39.81       0   90.55
Permanent Ineff=
       F       F
Bank Sta=33.38,47.63
XS Rating Curve= 0 ,0
Exp/Cntr=0.5,0.3

Type RM Length L Ch R = 1 ,1605.59 ,22.78,23.54,25
Node Photo=..\..\..\..\Corner Brook\Windshield Survey\CB photos\P1000703.JPG
XS GIS Cut Line= 5
344123.5905151375422913.68847656344142.2462768555422885.46252441
344137.1588745125422860.46691895344135.7728881845422849.03912354
 344138.025329595422843.67150879
#Sta/Elev= 19
       0      94     3.2   93.08    8.42   92.88    9.29   92.71    11.6   91.59
      13   89.94   18.32    85.2   21.06   82.36   23.96   82.16   29.14    81.8
   30.37   81.49   31.08   81.78   33.83   82.12   42.83   87.11   44.03   87.93
   52.64   90.04   60.74   91.65   70.91   95.94   76.67    96.2
#Mann= 3 , 0 , 0
       0     .06       0   23.96    .035       0   31.08    .055       0
Bank Sta=23.96,31.08
XS Rating Curve= 0 ,0
Exp/Cntr=0.3,0.1

River Reach=BellsB          ,M001

Type RM Length L Ch R = 1 ,1582.05 ,17.81,18.37,19.1
XS GIS Cut Line= 3
344135.5728759775422930.68328857344167.2293090825422893.19610596
344184.8796997075422881.19189453
#Sta/Elev= 26
       0   91.81    4.82   91.81       6   91.78    6.57   91.77    6.77   91.75
    7.32   91.72   16.69   91.18   24.35   84.37   26.89   82.57   29.01   81.61
   29.11   81.53   29.37    81.4   30.17  80.928   30.42   80.78   30.93   80.74
   32.27   80.41   36.11   80.99    36.7   81.05   37.07   81.11   49.07   87.64
   50.28   88.27   57.24   91.32   57.95   91.53   59.68   91.99   61.34   92.03
   70.41   92.03
#Mann= 3 , 0 , 0
       0     .06       0   30.17    .035       0   36.11     .05       0
Bank Sta=30.17,36.11
XS Rating Curve= 0 ,0
Exp/Cntr=0.3,0.1

Type RM Length L Ch R = 1 ,1563.67 ,18.98,19.42,20.26
XS GIS Cut Line= 2
344154.485717773 5422932.4967041344188.6195068365422900.46429443
#Sta/Elev= 17
       0   90.37     4.4    89.9    4.94   89.77    5.02   89.72    7.94    87.6
   16.04   81.55   18.95   80.51   19.66   80.26   19.87   80.19   21.39   79.96
   23.03    80.2   25.03   80.43   26.66   80.61   31.52   84.51   33.69   86.04
   38.24   89.37   46.81    91.5
#Mann= 3 , 0 , 0
       0     .06       0   19.66    .035       0   25.03     .05       0
Bank Sta=19.66,25.03
XS Rating Curve= 0 ,0
Exp/Cntr=0.3,0.1

Type RM Length L Ch R = 1 ,1544.26 ,15.64,15.21,13.49
XS GIS Cut Line= 3
344156.2185058595422952.52209473344191.1436767585422926.21228027
344193.3801269535422900.07452393
#Sta/Elev= 24
       0   89.87     9.3   88.46   12.68   88.33   13.01   88.19   13.72   87.61
   14.72   86.61    21.7   82.94    24.9   81.47   29.17   79.68   30.17   79.46
   31.18   79.04   34.26   79.66   34.58    79.7   35.43   80.42   36.69   81.77
   40.69   85.68   41.98   86.17   44.26   86.03   51.57   87.71   57.19   89.21
   64.21   91.23   66.31   91.45   66.89   91.58   69.96   91.64
#Mann= 3 , 0 , 0
       0     .06       0   30.17    .035       0   34.26     .05       0
Bank Sta=30.17,34.26
XS Rating Curve= 0 ,0
Exp/Cntr=0.3,0.1

Type RM Length L Ch R = 1 ,1529.04 ,18.66,13.38,5.34
XS GIS Cut Line= 5
344164.751708984 5422964.4151001344185.5438842775422946.23449707
344190.568725586 5422942.2520752344191.6082763675422933.94091797
344195.2468872075422900.35009766
#Sta/Elev= 25
       0   89.12    11.3   88.67   14.32   87.41   18.96   82.81   20.99   80.94
   22.42   78.71   22.69   78.63    23.5   78.38   26.26   78.24   27.62   78.42
   28.34   78.41   30.46   79.54   34.03   82.04   35.79    82.9   36.86    83.3
   39.89   84.83    41.9   85.66    43.7   85.68   47.51   86.61   51.11   86.07
    58.3    87.7   62.37   88.78   72.08   91.57   72.64   91.53   76.19   91.67
#Mann= 3 , 0 , 0
       0     .06       0   22.69    .035       0   28.34     .05       0
Bank Sta=22.69,28.34
XS Rating Curve= 0 ,0
Exp/Cntr=0.3,0.1

Type RM Length L Ch R = 1 ,1515.66 ,11.06,13.23,17.9
XS GIS Cut Line= 6
344184.1577148445422978.26690674344194.2072753915422968.57067871
 344196.113281255422958.70111084344192.9945068365422944.50292969
344192.4744873055422933.94091797344196.8062744145422900.52331543
#Sta/Elev= 30
       0   89.35    2.36   89.25    6.06   89.47      11    88.9   12.23   88.92
   13.45   88.64   13.96   88.37   21.44    82.8   22.08    82.4   26.35   78.59
   26.95   78.26   27.29   78.07   30.56    77.3   31.46   77.59    31.9   77.95
   35.55   80.82   36.48   81.01   36.73   80.96   42.33   82.67    43.3   83.43
   43.45   83.25   43.73   83.56   45.88   84.19   48.59   86.15   51.22   86.16
   53.64   86.77   58.16   86.11   65.27   87.69   78.87    91.5   82.83    91.7
#Mann= 3 , 0 , 0
       0     .06       0   26.95     .04       0    31.9     .05       0
Bank Sta=26.95,31.9
XS Rating Curve= 0 ,0
Exp/Cntr=0.3,0.1

Type RM Length L Ch R = 1 ,1502.43 ,17.13,18.96,22.01
XS GIS Cut Line= 3
344186.5355224615422980.11029053344206.0902709965422961.16369629
 344214.271301275422906.71710205
#Sta/Elev= 30
       0   89.38    1.43   89.32    4.08   89.44    5.57   89.05    9.53    88.6
   13.72   88.68   17.83   87.72   19.14   87.03   20.37   85.81   25.16   81.62
   27.31   79.42   28.97    77.1   29.69   76.43   30.31   75.02   31.57   72.94
   32.64    70.6   33.78   70.33   37.88   69.64   43.13   69.94   44.16   70.15
   48.73    71.1   49.41    71.1   50.21   71.64   53.59   72.89   54.25   73.26
   60.67   76.23   61.81   76.96   73.88   86.47   77.51   89.17   82.29   90.04
#Mann= 3 , 0 , 0
       0     .06       0   33.78     .04       0   44.16     .05       0
Bank Sta=33.78,44.16
XS Rating Curve= 0 ,0
Exp/Cntr=0.3,0.1

Type RM Length L Ch R = 1 ,1483.47 ,29.95,28.73,27.26
XS GIS Cut Line= 3
344212.0538940435422983.46130371344227.8212890635422952.29467773
344236.1381225595422917.14550781
#Sta/Elev= 29
       0   88.17     3.3   88.08    3.38   88.07    4.95   87.74    9.48   85.96
   10.07   85.74   10.18   85.64   11.42   84.71   17.49   78.35   18.26   77.46
   20.88   73.46   21.32   72.88   23.13   69.64    25.9   69.54   27.62   69.48
   31.82   69.16   32.71   68.89   34.93    69.2   37.64   69.34   38.28   69.38
   40.94   70.69   43.21   71.29   47.06   71.91      49   72.98   62.79   82.44
   66.97   85.97   67.43   86.29   69.07   87.22   71.05   88.13
#Mann= 3 , 0 , 0
       0     .06       0   27.62     .04       0   34.93     .05       0
Bank Sta=27.62,34.93
XS Rating Curve= 0 ,0
Exp/Cntr=0.3,0.1

Type RM Length L Ch R = 1 ,1454.75 ,46.23,48.12,48.46
XS GIS Cut Line= 3
344244.5089111335423006.18249512 344253.685485845422957.21392822
344267.0140991215422931.34307861
#Sta/Elev= 24
       0   86.22    6.43   85.78    9.67    85.8   16.53   86.26   19.97   86.07
   21.63   85.93   27.21   84.11   28.46    83.4   30.37    79.9   31.12   78.08
   32.64   74.06   33.21   72.45   35.11   68.66   36.75   68.27   37.85   68.26
   39.68   68.03   41.66   68.36   44.47   68.43   49.34   69.04   51.76   69.92
   67.78   81.67   71.24   83.88   73.64   85.83   78.92      87
#Mann= 3 , 0 , 0
       0     .06       0   37.85     .04       0   41.66     .05       0
Bank Sta=37.85,41.66
XS Rating Curve= 0 ,0
Exp/Cntr=0.3,0.1

Type RM Length L Ch R = 1 ,1406.62 ,45.67,48.12,50.82
XS GIS Cut Line= 4
 344270.56427002 5423014.0925293344285.178710938 5423009.6060791
344297.3618774415422973.44549561344310.1868896485422950.69970703
#Sta/Elev= 30
       0   83.57     .99   83.27   13.28   80.78   15.29   80.43   17.74   80.22
   18.94   79.99   20.99   79.62   23.43   78.97   24.17   78.46   26.07   76.73
   27.57   75.37   28.52   73.69   31.11   69.92   35.58   67.45   35.95    67.1
    36.8   66.91   37.65   66.49   40.58   67.04   41.19   67.11   41.46   67.12
   43.19   67.26   51.56   72.88   53.45   74.35   58.05   78.02   61.12   80.31
   69.81   85.96   70.74   86.67   74.53   87.63   75.64   87.75   79.56    88.1
#Mann= 3 , 0 , 0
       0     .06       0    36.8     .04       0   40.58     .05       0
Bank Sta=36.8,40.58
XS Rating Curve= 0 ,0
Exp/Cntr=0.3,0.1

Type RM Length L Ch R = 1 ,1358.51 ,45.41,48.12,49.91
XS GIS Cut Line= 2
344296.0416870125423047.56292725344356.4254760745422995.08648682
#Sta/Elev= 24
       0   81.66     .22   81.57    3.74   80.39   11.19   79.12   17.57   77.16
   18.22      77   21.35   74.77   27.13    70.7      28   70.14   34.76   66.21
   35.19   66.04   37.73   65.56   41.17   65.17   43.44   65.99   43.61   66.04
   45.52   66.38   47.76   68.24   57.26   75.62   58.22   76.05   69.36   78.79
   74.13   80.14    74.5   80.21   77.15   81.54      80   82.27
#Mann= 3 , 0 , 0
       0     .06       0   37.73     .04       0   43.44     .05       0
Bank Sta=37.73,43.44
XS Rating Curve= 0 ,0
Exp/Cntr=0.3,0.1

Type RM Length L Ch R = 1 ,1310.38 ,22.48,24.05,23.98
XS GIS Cut Line= 3
344324.8247070315423073.56048584344385.9348754885423040.35491943
344397.3156738285423038.21850586
#Sta/Elev= 29
       0   78.77    3.06   78.19    3.29   78.11   14.27   70.77   16.82   68.95
      19    67.8   23.13   66.31   25.02   65.92   27.33   65.54   30.99   65.09
      37   64.38   40.17    63.8   43.07   64.25   43.87   64.32   45.53    65.2
   48.38   66.55   48.95   66.99   50.99   68.27   52.08   69.16   52.17    69.2
   59.67   72.17   68.49   75.74   69.55   76.62   69.93   76.94   75.91   80.28
   77.69   81.24   77.86    81.3   79.55   81.65   81.13    81.8
#Mann= 3 , 0 , 0
       0     .06       0      37     .04       0   43.07     .05       0
Bank Sta=37,43.07
XS Rating Curve= 0 ,0
Exp/Cntr=0.3,0.1

Type RM Length L Ch R = 1 ,1286.33 ,28.88,24.08,12.48
XS GIS Cut Line= 5
344346.5858764655423091.49310303344359.7540893555423079.89208984
344375.348327637 5423074.5244751344384.5314941415423054.78552246
344395.6204833985423045.60870361
#Sta/Elev= 27
       0   78.89    5.63   77.47    8.18   76.37   11.07   73.16   12.18   71.46
   14.36    67.9   17.24    66.5   17.55   66.27   20.08   64.47   23.22   63.78
   24.56   63.46   26.31   63.04    26.8   62.81   27.39   63.01   28.94   63.28
   29.56   63.31   34.04   63.53   40.75   64.22   41.07   64.26   41.67   64.32
   44.89   66.29   55.53    70.2   55.81   70.42   62.21   75.81   63.35   76.68
      64   77.01   70.21   79.99
#Mann= 3 , 0 , 0
       0     .06       0   24.56     .04       0   29.56     .05       0
Bank Sta=24.56,29.56
XS Rating Curve= 0 ,0
Exp/Cntr=0.3,0.1

Type RM Length L Ch R = 1 ,1262.25 ,11.71,10.67,8.64
XS GIS Cut Line= 3
344373.4210815435423128.46972656344390.2106933595423060.81689453
344396.6876831055423048.99932861
#Sta/Elev= 24
       0    81.1    2.46   81.06   11.82   80.41   15.28   79.37    17.4   78.37
   19.73   77.08   23.73   73.96   25.09   72.28   26.62   70.51   29.39   65.75
   30.78   62.83   31.42    62.6   32.18   62.09   32.31    62.3   34.59    62.7
   42.46   63.81   42.98   63.99   57.64    63.9   58.75   64.02   66.88      69
   68.02   69.39   70.35   71.08   82.66   79.11   83.18   79.34
#Mann= 3 , 0 , 0
       0     .06       0   31.42     .04       0   34.59     .05       0
Bank Sta=31.42,34.59
XS Rating Curve= 0 ,0
Exp/Cntr=0.3,0.1

Type RM Length L Ch R = 1 ,1251.58 ,16.36,16.82,15.21
XS GIS Cut Line= 4
344386.2640991215423118.67730713344392.3284912115423104.82550049
344392.1552734385423087.51068115344403.0711059575423052.18829346
#Sta/Elev= 27
       0   78.98    1.27   78.29    3.91   76.54    5.31   75.26    8.12   71.37
   11.52   67.19   14.08   65.26   14.19   65.21   14.33   65.17   15.12   64.71
   18.38   63.04   19.27   62.49   19.53   62.41   20.51   62.26   24.03  61.741
   25.18   61.46   25.71   61.65   26.46   61.78   31.09   63.38   32.44   63.39
   34.72   63.37   46.38   63.65   47.27   63.93   47.36   63.94   48.22   64.47
   59.95   72.64   69.41   79.25
#Mann= 3 , 0 , 0
       0     .06       0   24.03     .04       0   26.46     .05       0
Bank Sta=24.03,26.46
XS Rating Curve= 0 ,0
Exp/Cntr=0.3,0.1

Type RM Length L Ch R = 1 ,1234.76 ,6.86,20.63,23.19
XS GIS Cut Line= 4
344395.1008911135423117.11907959344408.6157226565423102.40148926
344408.6157226565423084.91333008344412.2542724615423056.51708984
#Sta/Elev= 27
       0   73.55     .92   72.77    1.96   71.65    6.24   65.75    6.41   65.55
    6.43   65.53     8.8   64.51   12.38   63.36   13.09   62.96   14.63   62.72
   19.98   61.66   23.71   60.99   24.93   60.78   25.42   60.57   26.76  61.098
   28.16   61.44   31.29   61.62   34.35   61.79   37.47   62.08   43.55   62.52
   49.17   65.78   49.76   65.99   52.53   67.85   63.56   76.35   64.04   76.68
   64.62   77.08    66.1    77.9
#Mann= 3 , 0 , 0
       0     .06       0   23.71     .04       0   26.76     .05       0
Bank Sta=23.71,26.76
XS Rating Curve= 0 ,0
Exp/Cntr=0.3,0.1

Type RM Length L Ch R = 1 ,1214.13 ,15.14,13.55,13.08
XS GIS Cut Line= 3
344397.2103271485423117.85131836344450.7780761725423071.59112549
344453.648925781 5423060.8928833
#Sta/Elev= 27
       0   72.62    1.41   71.41    1.91   71.05    4.58   67.41     4.8   67.15
    7.92      65    8.39   64.68   12.07   63.56   13.04    63.1   24.19   61.01
   28.06   60.12   31.45   60.02   34.11   59.93   39.34   59.55   41.92   60.24
   42.35   60.32   43.05   60.58   44.72   62.02    45.8   62.84   46.96   63.85
   62.78   75.87   66.65   78.75   66.92   78.84   68.74   79.13   70.78   79.22
   71.26   79.25   81.85   80.38
#Mann= 3 , 0 , 0
       0     .06       0   34.11     .04       0   41.92     .05       0
Bank Sta=34.11,41.92
XS Rating Curve= 0 ,0
Exp/Cntr=0.3,0.1

Type RM Length L Ch R = 1 ,1200.58 ,17.09,17.6,17.74
XS GIS Cut Line= 2
344411.0806884775423127.57507324344455.4373168955423082.21032715
#Sta/Elev= 21
       0      71    6.14   66.79    6.66   66.45    9.87   65.27   11.64   64.61
   13.48    63.9   14.28   63.37   23.37   61.46   32.31   59.35    33.2   59.14
   34.93    58.9   36.39   59.54    36.9   59.72   39.18    60.5    39.3   60.53
   39.37   60.58    49.2   67.86   55.77   72.31   57.53   73.62   61.02    76.2
   63.45   77.88
#Mann= 3 , 0 , 0
       0     .06       0   32.31     .04       0    36.9     .05       0
Bank Sta=32.31,36.9
XS Rating Curve= 0 ,0
Exp/Cntr=0.3,0.1

Type RM Length L Ch R = 1 ,1182.98 ,17.91,16.97,16.65
XS GIS Cut Line= 3
344423.7293090825423137.27148438344451.4520874025423111.64550781
344464.7937011725423091.56030273
#Sta/Elev= 19
       0   72.88     .27   72.75    3.83   70.16    6.97   68.27    9.54   66.38
    13.4   63.45   15.34   62.34   25.65    60.4   31.25   59.27   33.78   58.59
   35.02   58.98   35.24   59.06   37.75   59.94   37.84   59.97      44   64.83
   47.57   67.31   51.05    69.3   59.62   75.23   61.86   76.83
#Mann= 3 , 0 , 0
       0     .06       0   31.25     .04       0   35.24     .05       0
Bank Sta=31.25,35.24
XS Rating Curve= 0 ,0
Exp/Cntr=0.3,0.1

Type RM Length L Ch R = 1 ,1166.01 ,11.83,12.83,13.49
XS GIS Cut Line= 3
344434.7974853525423155.41571045344474.6513061525423110.34112549
344474.8782958985423092.27392578
#Sta/Elev= 29
       0   74.51     .63   74.34    7.31    72.7   10.15   71.37   11.57   70.81
   11.82    70.7   14.11   68.03   15.34   66.94   20.02   63.39    21.9   62.05
      25   60.24   25.33   60.08   25.77   60.15   28.03   59.73   37.46   58.84
   40.29   58.57   42.21   58.39   42.81   58.78   44.66   59.34    45.1   59.53
   50.41    62.8   57.98   68.53   60.17   69.39      61   69.73   71.68   75.77
   71.77   75.79   72.05   75.88   73.99   76.19   78.24   76.81
#Mann= 3 , 0 , 0
       0     .06       0   37.46     .04       0   42.81     .05       0
Bank Sta=37.46,42.81
XS Rating Curve= 0 ,0
Exp/Cntr=0.3,0.1

Type RM Length L Ch R = 1 ,1153.18 ,11.32,11.3,11.26
XS GIS Cut Line= 3
344448.679870605 5423154.2401123344475.5363159185423129.82611084
344483.6798706055423115.62792969
#Sta/Elev= 21
       0   71.25    1.08   70.75    9.42   63.14     9.7   62.89   10.27   62.45
    10.5   62.34   15.88   59.27   20.47   58.93   25.39   58.95   25.46   58.95
   28.81   58.16   29.91    57.7   30.96   58.11   33.72   58.47   36.29   60.05
   36.84   60.38   40.91   61.57   46.43   65.54   47.97   66.12    50.2   67.43
   52.66   68.46
#Mann= 3 , 0 , 0
       0     .06       0   28.81     .04       0   30.96     .05       0
Bank Sta=28.81,30.96
XS Rating Curve= 0 ,0
Exp/Cntr=0.3,0.1

Type RM Length L Ch R = 1 ,1141.88 ,13.01,13.54,14.12
XS GIS Cut Line= 2
344458.3828735355423160.81970215344496.1552734385423126.18988037
#Sta/Elev= 24
       0    70.2     .88   70.17    3.52   69.42    5.89   68.62    6.48   67.83
    8.86   64.54   11.86   61.07    13.6   59.56   13.81   59.43   14.11   59.22
   15.36   58.79    22.1   57.32   23.95   56.72   26.11      57   27.88   57.23
    30.8   57.62   31.36    57.8   31.84   57.93   34.83   59.73   35.46   59.94
   48.05   64.99   49.73   65.42   50.94   65.93   51.24   66.04
#Mann= 3 , 0 , 0
       0     .06       0    22.1     .04       0   27.88     .05       0
Bank Sta=22.1,27.88
XS Rating Curve= 0 ,0
Exp/Cntr=0.3,0.1

Type RM Length L Ch R = 1 ,1128.34 ,10.91,10.45,10
XS GIS Cut Line= 4
344467.3927001955423166.01409912344472.4174804695423164.97528076
344476.5759277345423161.16607666344505.8582763675423138.31048584
#Sta/Elev= 21
       0   67.97    2.83   67.39    5.13   66.67    6.32   66.09    8.94    62.4
    9.25   62.13   10.77   60.82   11.57   60.13    15.2   58.43   18.58    56.9
   19.08   56.53   20.57   56.77   22.01  56.802   25.08   56.87   26.58   56.91
   27.02   56.93   29.77   57.01    41.2   61.41   41.44    61.5   43.95   62.56
   47.92    64.8
#Mann= 3 , 0 , 0
       0     .06       0   18.58     .04       0   22.01     .05       0
Bank Sta=18.58,22.01
XS Rating Curve= 0 ,0
Exp/Cntr=0.3,0.1

Type RM Length L Ch R = 1 ,1117.89 ,21.15,21.85,22.43
XS GIS Cut Line= 3
344466.2083129885423171.84667969344479.6917114265423173.35028076
344522.9801025395423135.09832764
#Sta/Elev= 28
       0   67.67    4.08   66.91    7.39   66.15    8.94   66.06   13.57   65.18
    14.8    65.1   15.17   64.94   21.02   59.24   21.77   58.51    22.1   58.39
   28.21   55.94   29.08   55.92    33.7   55.83   36.03   55.58   36.43  55.903
   40.23   57.13   40.43   57.26    46.2   60.51   50.11   62.74   53.02   64.34
    53.2   64.46   53.27    64.5   54.18   64.86   60.25    65.8    60.8   65.92
   65.94   67.89   68.16   68.89   71.33   69.44
#Mann= 3 , 0 , 0
       0     .06       0    33.7     .04       0   36.43     .05       0
Bank Sta=33.7,36.43
XS Rating Curve= 0 ,0
Exp/Cntr=0.3,0.1

Type RM Length L Ch R = 1 ,1096.03 ,13.27,18.23,17.07
XS GIS Cut Line= 4
344487.350524902 5423190.1350708344499.8256835945423183.20928955
344512.4743041995423174.37872314344529.1080932625423156.89068604
#Sta/Elev= 19
       0   63.34     2.7   62.35    6.71   59.39    6.89   59.29    7.85    58.7
   12.58   56.71   14.04   56.17   14.27   56.14   21.09   55.22   22.83   54.99
   23.94   54.61   24.73   54.89   26.51   55.14   28.17   55.36   29.69    56.3
   33.24   58.44      41   63.88   45.31   64.26   53.83   65.53
#Mann= 3 , 0 , 0
       0     .06       0   21.09     .04       0   26.51     .05       0
Bank Sta=21.09,26.51
XS Rating Curve= 0 ,0
Exp/Cntr=0.3,0.1

Type RM Length L Ch R = 1 ,1077.81 ,12.22,8.04,9.07
XS GIS Cut Line= 5
344497.9199218755423195.84912109344509.3555297855423189.44268799
344517.4990844735423191.86669922344525.1229248055423186.32592773
344533.7863159185423171.43511963
#Sta/Elev= 22
       0   60.62    8.56   55.97     8.8   55.84    9.27   55.81   13.11   55.47
   15.09    55.4   16.59   55.26   17.89   55.08    21.6   54.62   24.29   54.51
   25.89   54.24   30.49   54.46   31.03   54.46   31.06   54.46   33.15   55.29
   35.85   57.57    37.8   59.19   37.81    59.2   37.83   59.21   37.85   59.22
   47.84   63.83   48.26   63.88
#Mann= 3 , 0 , 0
       0     .06       0   24.29     .04       0   30.49     .05       0
Bank Sta=24.29,30.49
XS Rating Curve= 0 ,0
Exp/Cntr=0.3,0.1

Type RM Length L Ch R = 1 ,1069.76 ,4.65,5.09,6.22
XS GIS Cut Line= 3
344498.2136840825423203.04608154 344516.359497075423202.18109131
344560.6187133795423171.40948486
#Sta/Elev= 27
       0    61.4     .75   61.28    4.13   60.51    5.73   59.81   18.17   54.26
    18.7   53.97   19.25   53.93      20    53.9   28.68   53.92   32.03    53.7
    34.8   53.94   35.53   53.94   37.09   54.54    37.5   54.66   40.37   56.32
   48.58   58.31   49.02   58.39   49.24   58.43   52.47   59.54   55.98   60.33
   58.16   61.13    61.9   62.22   68.33   65.29    68.4   65.29   68.63   65.34
   70.71   65.45   72.07   65.53
#Mann= 3 , 0 , 0
       0     .06       0   28.68     .04       0    34.8     .05       0
Bank Sta=28.68,34.8
XS Rating Curve= 0 ,0
Exp/Cntr=0.3,0.1

Type RM Length L Ch R = 1 ,1064.67 ,7.87,13.03,14.53
XS GIS Cut Line= 4
344500.8823242195423206.66711426344519.248718262 5423205.6282959
344529.6447143555423198.87548828344557.5408935555423186.75512695
#Sta/Elev= 20
       0   60.67     .51   60.56    3.25   59.77    3.37   59.71   15.92   53.91
   17.59   53.47   18.05   53.42    18.4    53.4   23.02   53.41   24.25   53.45
   28.36   53.49   30.79   53.19   34.57   53.48   35.28   53.47   39.41   55.71
   41.08   56.68    42.6   56.96   52.11   58.71   52.46   58.76   61.21   60.91
#Mann= 3 , 0 , 0
       0     .06       0   28.36     .04       0   34.57     .05       0
Bank Sta=28.36,34.57
XS Rating Curve= 0 ,0
Exp/Cntr=0.3,0.1

Type RM Length L Ch R = 1 ,1051.64 ,18.34,19.28,20.15
XS GIS Cut Line= 5
344501.2288818365423211.86169434344520.6348876955423212.72729492
344535.882324219 5423210.6494751344552.8624877935423207.01348877
344560.8328857425423202.33850098
#Sta/Elev= 21
       0   60.15    4.02   58.95    4.36    58.8   13.42   54.56   19.43   52.97
    20.1   52.79   21.93   52.61    29.3   52.29   29.74   52.27   34.81   51.97
    35.5   52.29   36.54   52.53   40.12    55.1   42.71   56.77   48.52   57.61
   52.18   58.17   55.78   58.73   56.13   58.81   57.46   59.13   59.47    60.5
   61.42   61.51
#Mann= 3 , 0 , 0
       0     .06       0    29.3     .04       0    35.5     .05       0
Bank Sta=29.3,35.5
XS Rating Curve= 0 ,0
Exp/Cntr=0.3,0.1

Type RM Length L Ch R = 1 ,1032.36 ,11.78,10.72,9.73
XS GIS Cut Line= 4
 344503.654479985423234.71728516344520.9813232425423230.90789795
344551.476501465 5423229.0032959344556.327880859  5423220.519104
#Sta/Elev= 19
       0   61.27     .12   61.24     .77   60.95    4.44   58.77    4.94   58.52
   10.45   54.69   17.74   52.66    20.8   51.78   21.31   51.69   26.13   51.54
   29.99   51.41   32.07   50.97   33.31    51.4   36.46   53.45   41.33   56.26
   42.55   56.58   45.54   56.67    48.3   56.89   58.07   57.92
#Mann= 3 , 0 , 0
       0     .06       0   29.99     .04       0   33.31     .05       0
Bank Sta=29.99,33.31
XS Rating Curve= 0 ,0
Exp/Cntr=0.3,0.1

Type RM Length L Ch R = 1 ,1021.64 ,9.54,7.54,5.22
XS GIS Cut Line= 3
344494.0515136725423248.73413086344549.3900756845423237.51171875
344568.1500854495423221.73791504
#Sta/Elev= 26
       0      65     .65   64.86    3.32    64.2   18.54    59.9   21.32   57.69
   30.29   51.53   33.56   51.04   37.02   50.69   41.48   50.03   43.33   50.63
   44.28   50.83   45.02   50.93    47.3   51.43   47.35   51.45   47.64   51.63
   52.52   54.25   56.15   56.41   56.47   56.47    56.6   56.48   57.16    56.7
   57.78   56.88   64.88   56.96   71.97   57.72   74.79   57.76   75.43   57.81
   80.98   58.42
#Mann= 3 , 0 , 0
       0     .06       0   37.02     .04       0   43.33     .05       0
Bank Sta=37.02,43.33
XS Rating Curve= 0 ,0
Exp/Cntr=0.3,0.1

Type RM Length L Ch R = 1 ,1014.11 ,8.95,7.86,6.39
XS GIS Cut Line= 4
344516.8228759775423257.22650146344540.9071044925423245.27929688
344550.4368896485423238.00708008344567.9368896485423222.94311523
#Sta/Elev= 26
       0   60.12     .67   59.93    4.16   57.09    5.09   56.58   11.73   51.73
   13.33   51.63   18.96   50.34   19.95   50.12   20.57   49.69   21.35   49.46
   24.27   49.99   24.42   50.02   25.13   50.18   26.88   50.48   30.33   51.12
   32.69   52.64   38.52   56.67   38.87   56.71   38.98   56.72   39.25   56.83
   39.56   56.91    47.3      57    53.2   57.63   55.61   57.67   56.15   57.71
   61.96   58.35
#Mann= 3 , 0 , 0
       0     .06       0   18.96     .04       0   24.42     .05       0
Bank Sta=18.96,24.42
XS Rating Curve= 0 ,0
Exp/Cntr=0.3,0.1

Type RM Length L Ch R = 1 ,1006.24 ,12.82,9.82,6.31
XS GIS Cut Line= 4
344522.0208740235423267.09588623344547.3181152345423249.26171875
344553.2091064455423236.96807861344568.2835083015423224.32830811
#Sta/Elev= 28
       0   59.82     .85   59.64    11.1   53.01   11.68   52.62   12.45   52.04
   15.95   51.81   16.66   51.74   16.76   51.73    20.1   49.43   20.18   49.36
   20.21   49.34   20.51   49.15   25.84   49.52   25.97   49.53   26.78   49.64
   29.69   50.16   30.95   50.15   31.96   50.24    33.5   50.55   41.89   56.34
   43.22   56.94   43.49   56.98   44.58   56.97   50.79   57.04   55.22   57.52
   56.97   57.54   57.37   57.57   64.26   58.34
#Mann= 3 , 0 , 0
       0     .06       0    20.1     .04       0   25.84     .05       0
Bank Sta=20.1,25.84
XS Rating Curve= 0 ,0
Exp/Cntr=0.3,0.1

Type RM Length L Ch R = 1 ,996.42  ,8.2,9.15,9.17
XS GIS Cut Line= 5
344531.2041015635423274.71447754344545.7587280275423265.53771973
344555.1151123055423247.70330811344565.1646728525423238.00708008
344569.3231201175423227.96447754
#Sta/Elev= 26
       0   58.24    5.26   53.59    7.26   52.01    7.82   51.82     9.4   51.16
   12.28   50.88    13.1   50.71   17.21   50.52   17.39   50.51   19.05   49.28
   19.44    49.3   21.36  48.595      22   48.36   22.12   48.11   25.24  48.554
   27.36   48.72   29.82   48.92   36.28   50.19   37.35   50.92   38.67   51.69
   42.36   52.78   48.71   56.55    50.3   56.73   51.31   56.78   53.91   56.96
   62.18    58.2
#Mann= 3 , 0 , 0
       0     .06       0   21.36     .04       0   25.24     .05       0
Bank Sta=21.36,25.24
XS Rating Curve= 0 ,0
Exp/Cntr=0.3,0.1

Type RM Length L Ch R = 1 ,987.27  ,17.06,13.75,13.19
XS GIS Cut Line= 4
 344535.189270025423279.56268311344554.0755004885423269.34692383
344558.7537231455423260.34307861344572.0952758795423234.54412842
#Sta/Elev= 24
       0   57.24     .52   57.08    1.25   56.25    7.51   50.81   19.32   50.37
   20.67   50.24   20.76   50.24   21.47    50.1   22.11   50.06   23.08    49.6
   26.65   48.16   27.99   47.62   28.63   47.51    29.1   47.46   30.53   47.17
   31.62    47.6   32.35   47.76   34.86   48.29   36.79   48.74   42.27   51.88
   49.63   56.09   50.82   56.25   58.13   56.72   60.66   57.09
#Mann= 3 , 0 , 0
       0     .06       0   27.99     .04       0   32.35     .05       0
Bank Sta=27.99,32.35
XS Rating Curve= 0 ,0
Exp/Cntr=0.3,0.1

Type RM Length L Ch R = 1 ,973.52  ,11.18,22.09,23.3
XS GIS Cut Line= 3
344553.4329223635423296.50427246344561.8582763675423291.50048828
344583.8804931645423229.90710449
#Sta/Elev= 28
       0      52      .5   51.14    1.42   50.62    4.04   49.73    4.18   49.68
    4.59   49.44    4.75   49.41    6.22   49.36    7.96   49.41     9.8    49.4
   10.28   49.41    11.4   49.42   17.95   49.17    31.1   47.79   33.04   47.41
    35.2   46.99   37.33   46.79   38.63   47.11   39.22   47.34   41.15   49.24
   48.66   54.37   48.94   54.56   50.03    55.2   52.27    55.3   65.34   56.25
   74.17    57.6   74.98   57.75   75.21   57.78
#Mann= 3 , 0 , 0
       0    .047       0   33.04    .037       0   39.22    .047       0
Bank Sta=33.04,39.22
XS Rating Curve= 0 ,0
Exp/Cntr=0.3,0.1

Type RM Length L Ch R = 1 ,951.43  ,14.71,19.93,24.34
XS GIS Cut Line= 6
344554.1068725595423297.98010254344563.1168823245423292.78552246
 344567.795104985423284.30133057344575.4188842775423284.30133057
344589.800109863  5423276.855896344605.0477294925423250.88372803
#Sta/Elev= 18
       0   51.12     4.7   49.37   12.74   49.38   16.71   49.22   25.29   48.18
   27.71   48.08   38.27   47.21   42.97   46.78   45.56   46.46   49.14   45.77
   49.21   45.96   50.68  46.402   55.76   48.11   61.13   52.81   67.89   54.94
   68.22   54.96   69.53   55.82    74.1    56.2
#Mann= 3 , 0 , 0
       0    .047       0   45.56    .037       0   50.68    .047       0
Bank Sta=45.56,50.68
XS Rating Curve= 0 ,0
Exp/Cntr=0.3,0.1

Type RM Length L Ch R = 1 ,931.51  ,6.29,6.11,6.81
XS GIS Cut Line= 6
344554.6267089845423299.19207764344563.9832763675423293.65130615
344584.6021118165423290.88092041344593.6121215825423291.40032959
344610.4188842775423287.41790771 344616.82989502  5423279.453125
#Sta/Elev= 26
       0    51.1    4.84   49.31   10.87   49.33   15.36   49.24   16.04   49.22
   16.57   49.06   17.29   48.95   21.53   48.38   31.73   46.97   31.84   46.96
   40.76   45.51   43.31   45.14   43.75   44.86   44.73   45.13   45.26   45.14
   48.89   45.26   50.33   46.05   51.26   46.56   52.32   47.04   55.62   49.37
   56.11   49.71   58.03   51.26   58.19   51.37   59.26   51.62   62.93    52.4
   68.25   52.99
#Mann= 3 , 0 , 0
       0    .047       0   43.31    .037       0   45.26    .047       0
Bank Sta=43.31,45.26
XS Rating Curve= 0 ,0
Exp/Cntr=0.3,0.1

Type RM Length L Ch R = 1 ,925.41  ,20.85,23.72,25.32
XS GIS Cut Line= 4
 344567.13067627 5423304.6663208344580.9411010745423298.03607178
344616.3770751955423294.27911377344625.477478027 5423285.9730835
#Sta/Elev= 23
       0    48.8     .89    48.8    7.38   48.77   10.72   47.66   15.32   47.14
   16.76   46.94   23.27   45.94   29.05   45.93   30.57  45.115   30.99   44.69
   32.18    44.7   33.01   45.09   33.27   45.15   38.03   45.44   38.22   45.62
   39.22   46.49   42.94   49.32   43.34   49.45   46.45   50.45   50.95   51.07
   53.06   51.47   56.17   52.12   63.28   52.88
#Mann= 3 , 0 , 0
       0    .047       0   30.57    .037       0   33.27    .047       0
Bank Sta=30.57,33.27
XS Rating Curve= 0 ,0
Exp/Cntr=0.3,0.1

Type RM Length L Ch R = 1 ,901.68  ,25.83,24.41,23.27
XS GIS Cut Line= 4
344564.8494873055423325.16430664344587.0278930665423317.02648926
344603.3148803715423320.48931885344607.9932861335423311.83190918
#Sta/Elev= 23
       0   51.03    7.77   48.12    8.46   47.85    9.65   47.83    9.84   47.82
      13   47.78   16.45   47.68   20.67   47.52   21.79   47.28   23.62   46.51
   26.66   44.93   28.09    44.2   28.92   44.06   31.46   43.69   33.23  44.103
   35.23   44.35   36.35   44.49   36.41   44.53   36.86   44.84   39.97   46.98
   40.28   47.22   42.99   47.94   50.12   48.39
#Mann= 3 , 0 , 0
       0    .047       0   28.92    .037       0   33.23    .047       0
Bank Sta=28.92,33.23
XS Rating Curve= 0 ,0
Exp/Cntr=0.3,0.1

Type RM Length L Ch R = 1 ,877.27  ,29.64,19.87,13.78
Node Photo=..\..\..\..\Corner Brook\Windshield Survey\CB photos\Google\2119 US.jpg
XS GIS Cut Line= 3
344554.6296997075423343.80212402344603.0496826175423343.29449463
344609.8696899415423314.36651611
#Sta/Elev= 24
       0   53.04   15.03   50.61   19.88   48.56   23.72   47.03   29.35   46.64
   31.18   46.44   34.88    43.8   34.89    43.8    34.9    43.8   37.51   43.61
   39.79   43.45   41.89   43.18   42.23   43.52   44.77   44.64   48.11    46.4
   48.42   46.43   52.04   46.69   55.35      47   56.08   47.02   56.85   47.06
   57.34    47.1   72.12   47.81   72.97   47.84   78.14    48.2
#Mann= 3 , 0 , 0
       0    .047       0   37.51    .037       0   42.23    .047       0
Bank Sta=37.51,42.23
XS Rating Curve= 0 ,0
Exp/Cntr=0.3,0.1

Type RM Length L Ch R = 1 ,857.41  ,43,43.13,43.22
Node Photo=..\..\..\..\Corner Brook\Windshield Survey\CB photos\P1000700.JPG
XS GIS Cut Line= 4
      344577.572      5423397.11      344604.327     5423352.442
      344604.327     5423352.442      344611.617      5423321.54
#Sta/Elev= 24
       0      50    1.36      49    2.71      48    3.32      47    4.12      46
   15.03      45   28.06   44.93   30.12      45   35.65      43   35.87   42.75
   36.66   42.61   38.69   42.57   39.26   42.16   39.88   42.16   40.89   42.54
   41.35  42.627   42.55  42.853    43.8   42.95   44.83      44   46.95      45
   47.78   45.43   50.63      46   66.44      47   83.82      48
#Mann= 3 , 0 , 0
       0    .047       0   35.87    .037       0   41.35    .047       0
#XS Ineff= 2 , 0
       0   35.52      45   40.77       0    45.4
Permanent Ineff=
       F       F
Bank Sta=35.87,41.35
XS Rating Curve= 0 ,0
Exp/Cntr=0.5,0.3

Type RM Length L Ch R = 2 ,840     ,,,
Node Photo=..\..\..\..\Corner Brook\Windshield Survey\CB photos\P1000697.JPG
BEGIN DESCRIPTION:
Wellington Street (Structure #2119)
END DESCRIPTION:
Bridge Culvert--1,0,-1,-1, 0
Deck Dist Width WeirC Skew NumUp NumDn MinLoCord MaxHiCord MaxSubmerge Is_Ogee
8.7,16,1.67,0, 16, 16, 44.76, , 0.98, 0, 1,0.3,,
       0     .83    5.55   12.75   17.14   20.65   25.29   29.78    36.4   42.14
   46.88   52.62    57.3   61.71   72.14   83.81
      45      45   44.83   44.89   44.76   45.04   45.08   45.17    45.4   45.49
   45.75   46.01   46.19    46.4      47      48
                                                                                
                                                
       0    8.83   13.32   17.31   22.94   27.33   30.84   35.48   39.97   46.59
   52.32   57.07   62.81   67.49    71.9      80
      45      45   44.82   44.69   44.89   44.76   45.04   45.08   45.17    45.4
   45.49   45.75   46.01   46.19    46.4      47
                                                                                
                                                
BR Coef=-1 , 0 , 0 ,, 0 ,,,0.8,-1,,0,
WSPro=,,,, 1 ,,,, 0 ,,,, 0 ,,,,-1 ,-1 ,-1 , 0 , 0 , 0 , 0 , 0
Culvert=1,1.8,,40,0.03,0.5,1,1,1,42.61,36.42,38.79,37.42,Culvert #2  , 0 ,2
Culvert Bottom n=0.03
Culvert=1,2.4,,35.7,0.03,0.5,1,1,1,42.18,39.57,39.94,39.88,Culvert #1  , 0 ,4.75
Culvert Bottom n=0.03
BC Design=,, 0 ,, 0 ,,,,,,
BC Use User HTab Curves=0
BC User HTab FreeFlow(D)= 0

Type RM Length L Ch R = 1 ,816.09  ,5.75,5.97,5.64
Node Photo=..\..\..\..\Corner Brook\Windshield Survey\CB photos\Google\2119 DS.jpg
XS GIS Cut Line= 2
 344595.072082525423433.64447021344636.2438964845423365.05230713
#Sta/Elev= 28
       0      46    5.81      46   20.37      45   27.28   44.56   28.35      44
   29.66   43.44   30.78   43.22   31.04      43   32.44      42   33.65      41
   34.63      40   35.38   39.99   36.47    39.6   36.58   39.34   36.71   39.12
   36.97    38.9   38.85   38.69   39.24   38.54   41.55  39.018   42.14   39.14
   42.24      40    42.9   40.49   43.35      41   43.96      42   45.36   42.72
   50.46      43   68.59      44      80      45
#Mann= 3 , 0 , 0
       0    .047       0   36.97     .04       0   41.55    .047       0
#XS Ineff= 2 , 0
       0   36.52    42.5   41.07       0    43.5
Permanent Ineff=
       F       F
Bank Sta=36.97,41.55
XS Rating Curve= 0 ,0
Exp/Cntr=0.5,0.3

Type RM Length L Ch R = 1 ,810.13  ,13.89,13.76,13.13
Node Photo=..\..\..\..\Corner Brook\Windshield Survey\CB photos\Google\2118 US.jpg
XS GIS Cut Line= 2
 344598.634704595423438.42871094 344639.806701665423369.83648682
#Sta/Elev= 21
       0   44.97    1.85   44.72    8.24      44   14.18      43   31.04      42
   34.79      41   35.57      40      36      39   36.23      38   37.14    37.8
   38.32   37.81    40.3      38   41.16   38.48   43.02      39   43.82   39.78
   44.01      40   45.03      41   53.19      42   61.49      43   78.46      44
      80   44.14
#Mann= 3 , 0 , 0
       0    .047       0      36     .04       0   43.02    .047       0
#XS Ineff= 2 , 0
       0   36.33   41.35   43.45       0   41.47
Permanent Ineff=
       F       F
Bank Sta=36,43.02
XS Rating Curve= 0 ,0
Exp/Cntr=0.5,0.3

Type RM Length L Ch R = 3 ,800     ,,,
Node Photo=..\..\..\..\Corner Brook\Windshield Survey\CB photos\P1000695.JPG
BEGIN DESCRIPTION:
Blackwood's Hill Road (Structure #2118)
END DESCRIPTION:
Bridge Culvert--1,0,-1,-1, 0
Deck Dist Width WeirC Skew NumUp NumDn MinLoCord MaxHiCord MaxSubmerge Is_Ogee
1.3,6.5,1.67,0, 19, 19, 40.3, , 0.98, 0, 0,0,,
       0    6.76    19.8   28.39   31.26   35.12   36.33   36.34   36.74   39.15
   43.44   43.84   43.85   43.92   47.96   51.45   58.47   70.99   80.01
      43      43      42   41.51   41.43   41.35   41.43   41.43   41.43   41.45
   41.47   41.47   41.47   41.47   41.52   41.64      42      43      44
                                                      35   39.28   39.68   39.68
   39.68   39.28      35
       0    4.96   18.86   30.87   33.96   37.05   37.06   37.46   38.61   43.43
   44.23   44.56   44.57   47.15   50.75    56.9   68.35   76.01      80
      43      43      42   41.73   41.43   41.43   41.43   41.43   41.43   41.45
   41.47   41.47   41.47   41.52   41.64      42      43      43   43.09
                                              35   39.28   39.68   39.68   39.68
   39.68   39.28      35
BR Coef=-1 , 0 , 0 ,, 0 ,,,0.8,-1,,0,
WSPro=,,,, 1 ,,,, 0 ,,,, 0 ,,,,-1 ,-1 ,-1 , 0 , 0 , 0 , 0 , 0
BC Design=,, 0 ,, 0 ,,,,,,
BC Use User HTab Curves=0
BC User HTab FreeFlow(D)= 0

Type RM Length L Ch R = 1 ,796.37  ,12.75,14.1,16.38
Node Photo=..\..\..\..\Corner Brook\Windshield Survey\CB photos\Google\2119 DS.jpg
XS GIS Cut Line= 2
344606.2000732425423449.90393066344647.3718872075423381.31170654
#Sta/Elev= 27
       0   43.61    7.03      43   10.37      42   30.95      41    32.9      40
   33.72      39   34.06      38   34.49      37   34.95      36   35.67  35.014
   35.68      35   37.11   34.57   37.91   34.33   39.01      35   39.67    35.3
   41.49      36   42.44  36.367   44.08      37   44.26  37.127   44.66  37.408
    45.5      38   47.57      39   49.02      40   50.25      41   62.63      42
   76.01      43   80.01   43.09
#Mann= 3 , 0 , 0
       0     .06       0   34.95     .04       0   41.49     .05       0
#XS Ineff= 2 , 0
       0   37.05   40.56   44.57       0   40.56
Permanent Ineff=
       F       F
Bank Sta=34.95,41.49
XS Rating Curve= 0 ,0
Exp/Cntr=0.5,0.3

Type RM Length L Ch R = 1 ,782.27  ,8.97,9.53,9.31
XS GIS Cut Line= 4
 344608.363281255423447.75390625344615.467102051 5423437.3651123
344627.9425048835423431.82427979344649.0811157235423417.27990723
#Sta/Elev= 25
       0   43.36    3.08   43.14    3.22   43.12    5.48   42.42    8.26   41.72
   12.59   40.81    13.4   40.46   13.46   40.42   14.12   40.33   14.38   40.31
   24.92   40.14   25.18   39.99   25.86   39.72   26.24   39.23   28.83   36.01
   29.96   34.47   29.98   34.46   30.82   33.92   32.94   34.07   36.58    34.3
   39.97   34.34   40.85   34.88   44.92   38.06    48.2   40.48   51.89   40.59
#Mann= 3 , 0 , 0
       0     .06       0   29.98     .04       0   36.58     .05       0
Bank Sta=29.98,36.58
XS Rating Curve= 0 ,0
Exp/Cntr=0.3,0.1

Type RM Length L Ch R = 1 ,772.73  ,5.73,5.99,6.14
XS GIS Cut Line= 5
344608.8828735355423447.75390625 344614.947326665423438.75030518
344622.0513305665423436.49932861 344631.234497075423440.30847168
 344654.798889165423424.72528076
#Sta/Elev= 28
       0   43.31    2.64   43.13    2.85   43.09    6.07    42.1    9.88   41.15
   10.86   40.94   11.26   40.76   12.87   40.17   18.31      40   19.11   39.93
   23.72   39.89   25.31   39.68   25.99   39.33   28.25   38.59   29.82   37.75
   30.09   37.68   31.22   36.53   33.68   32.84   33.71   32.84   42.78   31.37
   43.72   31.21   44.19   30.94   44.25   31.18   44.48  31.431   50.56   38.07
   53.38   39.54    53.9   39.59    56.5   39.69
#Mann= 3 , 0 , 0
       0     .06       0   42.78     .04       0   44.48     .05       0
Bank Sta=42.78,44.48
XS Rating Curve= 0 ,0
Exp/Cntr=0.3,0.1

Type RM Length L Ch R = 1 ,766.74  ,6.37,6.42,6.54
XS GIS Cut Line= 6
 344609.576110845423449.13909912344616.6801147465423445.50311279
344631.581115723 5423445.8493042344636.6058959965423443.42529297
344655.1455078135423432.17071533344657.5712890635423427.84191895
#Sta/Elev= 30
       0   43.27    2.82      43    3.31   42.89    3.52   42.79    7.98   40.76
   10.35   39.62   15.66   39.42   16.45   39.32   22.89   38.62   25.39   38.49
   26.02   38.24   26.78   37.84   27.51   36.74   28.46   35.24      30   32.84
    32.3   32.35   37.19   31.31   38.19  31.075   38.89   30.91   39.28   30.65
   39.66    31.1   42.13   32.74   44.32   34.06    44.7   34.47   49.79   37.07
   50.15   37.26   50.22   37.29   52.99   38.96   53.08   38.98   55.11   39.17
#Mann= 3 , 0 , 0
       0     .06       0   38.19     .04       0   39.66     .05       0
Bank Sta=38.19,39.66
XS Rating Curve= 0 ,0
Exp/Cntr=0.3,0.1
