HEC-RAS study Corner_Brook2.prj: Corner_Brook2

--- Corner_Brook2.g02 (geometry) --- (continued)

Type RM Length L Ch R = 1 ,828.33  ,50.77,43.78,31.08
XS GIS Cut Line= 4
      345164.294     5423647.316      345168.009     5423651.144
      345249.904     5423738.293      345378.862     5423831.031
#Sta/Elev= 20
       0       6    5.33    5.83   34.89    3.74   41.92    3.62   48.13    2.46
   54.75    1.29   55.06    1.26   58.59     .77   60.77    1.01   70.65    1.35
   73.94    1.44   94.38       2  103.58    2.17  124.92    2.21  212.31    2.46
  225.59    2.55  247.57    4.18  248.51    4.31   278.1       5  283.77       6
#Mann= 3 , 0 , 0
       0    .055       0   54.75    .035       0   70.65    .055       0
Bank Sta=54.75,70.65
XS Rating Curve= 0 ,0
Exp/Cntr=0.3,0.1

Type RM Length L Ch R = 1 ,784.55  ,56.66,44.7,40.93
XS GIS Cut Line= 5
      345140.972     5423686.402       345141.44     5423687.378
      345158.944     5423719.864      345265.845     5423765.156
      345371.196     5423846.325
#Sta/Elev= 22
       0       6    1.08    5.79    1.41    5.77   14.55    3.66   15.48    3.56
   28.65    3.08   37.98    2.97   50.24    2.91   55.27    2.09   58.77    1.47
   61.54     .82   71.65    1.27   77.13    1.42  107.56    2.06  154.08    2.23
  194.93    2.34  219.57    2.52  245.66    4.48   253.7    4.66  257.47     4.7
  276.33       5  287.08       6
#Mann= 3 , 0 , 0
       0    .045       0   58.77    .035       0   71.65    .045       0
Bank Sta=58.77,71.65
XS Rating Curve= 0 ,0
Exp/Cntr=0.3,0.1

Type RM Length L Ch R = 1 ,739.85  ,37.83,43.49,53.15
XS GIS Cut Line= 4
      345076.712     5423735.284      345137.039     5423763.084
      345236.439     5423792.134      345351.066      5423879.91
#Sta/Elev= 22
       0       6     .02    5.91    5.71    3.38    6.21    3.18    6.96    3.19
   50.21    3.36   66.42    3.23   70.74    3.19   88.31    2.08   89.02    1.93
    90.8   1.558   93.38     .82     110    1.39  119.17     1.6  137.07    1.89
  169.98    2.03  170.06    2.03  226.25    2.44  240.15    3.48  272.74     4.2
  303.67       5  314.36       6
#Mann= 3 , 0 , 0
       0    .045       0    90.8    .035       0  119.17    .045       0
Bank Sta=90.8,119.17
XS Rating Curve= 0 ,0
Exp/Cntr=0.3,0.1

Type RM Length L Ch R = 1 ,696.36  ,64.23,36.99,20.23
XS GIS Cut Line= 4
      345063.287     5423758.789      345096.278     5423783.749
      345132.515     5423802.491      345321.259     5423898.327
#Sta/Elev= 24
       0       6    3.63       5    5.14       4   41.37    3.52   43.54    3.54
   55.45    3.68    61.4    3.57   90.68    1.66   95.01    1.38   98.76     .64
  110.67     .88  117.99    1.36  122.44    1.66  132.24    2.74  188.88    2.27
  192.82    2.43  200.02    2.34  200.92    2.36  217.79    2.75  269.67    3.97
  269.99    3.98  273.09    4.45  279.33       5  293.85       6
#Mann= 3 , 0 , 0
       0    .045       0   95.01    .035       0  117.99    .045       0
Bank Sta=95.01,117.99
XS Rating Curve= 0 ,0
Exp/Cntr=0.3,0.1

River Reach=CornerB         ,M001

Type RM Length L Ch R = 1 ,659.37  ,6.01,15.44,16.77
XS GIS Cut Line= 6
      345019.923     5423888.005      345062.738     5423875.777
      345130.858       5423844.8      345159.361     5423841.647
      345204.919     5423855.768      345306.953     5423901.466
#Sta/Elev= 23
       0       6   52.88    4.49   81.27    3.51   82.46    3.57   91.21    3.35
  104.43    3.36  105.52    3.24  110.73   1.506   112.4     .95  118.32     .88
  120.42     .75  123.84     .86  125.39    1.28   141.4     1.5  148.29    2.13
  173.91    1.99  194.51    2.71  225.58    2.34  289.42    3.83  290.06    3.85
  293.74    4.37  295.96       5  307.62       6
#Mann= 3 , 0 , 0
       0    .045       0  110.73    .035       0   141.4    .045       0
Bank Sta=110.73,141.4
XS Rating Curve= 0 ,0
Exp/Cntr=0.3,0.1

Type RM Length L Ch R = 1 ,608.52  ,41.15,38.4,36.15
XS GIS Cut Line= 6
      345020.472     5423889.988      345061.819     5423890.967
      345102.693     5423890.907      345177.941      5423897.73
      345254.053     5423918.189      345265.011     5423928.885
#Sta/Elev= 23
       0       6   41.36    5.04   45.94       5   49.74    4.79    67.8    4.29
   78.37    3.64   87.72    3.42   89.41    2.52      91     2.6   95.94    2.08
   98.56   1.668   103.7     .76  107.68    1.15  114.64   1.652  127.39    2.56
  140.25    2.74  197.16    2.33  208.45    3.77   210.4     3.8  223.29       3
   236.6    3.36  237.21       4  251.92       5
#Mann= 3 , 0 , 0
       0    .045       0   98.56    .035       0  114.64    .045       0
Bank Sta=98.56,114.64
XS Rating Curve= 0 ,0
Exp/Cntr=0.3,0.1

Type RM Length L Ch R = 1 ,570.12  ,24.66,34.29,42.16
XS GIS Cut Line= 3
      345060.639     5423923.096      345070.954     5423931.842
      345264.424     5423933.617
#Sta/Elev= 29
       0       6    6.11    4.91   12.82    4.48   17.49     3.6   19.63    3.56
   40.62    2.34    58.1    2.64   59.04    2.61    69.2    1.28    73.2     .61
   78.27    1.11   81.71   1.277   92.91    1.82   94.33    1.89   95.97    1.93
   99.84    2.22  101.05    2.23  106.61    2.53  110.05    2.46  129.57    2.36
  143.11    2.38  154.45    2.42  163.57    2.43  188.48    3.04  189.63    3.07
  200.02    3.38  200.77    3.41   203.1    4.24     207       5
#Mann= 3 , 0 , 0
       0    .045       0    69.2    .035       0   81.71    .045       0
Bank Sta=69.2,81.71
XS Rating Curve= 0 ,0
Exp/Cntr=0.3,0.1

Type RM Length L Ch R = 1 ,535.83  ,15.48,15.61,15.92
XS GIS Cut Line= 6
      345041.667     5423921.564      345048.939     5423951.247
      345097.825      5423955.91      345179.627     5423978.872
      345254.305     5423970.477      345277.023      5423969.84
#Sta/Elev= 23
       0       6    5.94       5   13.47       4   24.91       3   44.79    3.21
   78.78    2.85   87.35    2.44    91.1    2.49  103.75     .84  104.68     .79
  108.59     .56  136.62     .56  137.63     .78  138.99      .9  144.57    2.32
  164.63    2.61  177.83    2.89  200.21    3.07  225.72    3.05  231.31    3.18
  235.59    3.99  239.78    4.34  262.51       5
#Mann= 3 , 0 , 0
       0    .045       0  104.68    .035       0  138.99    .045       0
#XS Ineff= 2 , 0
       0    54.3       5               0
Permanent Ineff=
       F       F
Bank Sta=104.68,138.99
XS Rating Curve= 0 ,0
Exp/Cntr=0.3,0.1

Type RM Length L Ch R = 1 ,520.22  ,48.43,48.15,48.46
XS GIS Cut Line= 6
      344948.158     5423933.212      344970.145     5423938.241
      344987.893     5423961.271      345093.136     5423970.747
      345200.729     5424001.107      345276.787     5423972.194
#Sta/Elev= 22
       0       6   32.75       5   34.12       4   38.38       3  108.19    2.54
  125.31    2.69  145.78    2.54  166.66    2.28  175.28    1.91  182.41    .966
  183.94      .8  185.21     .55  212.24     .55  212.62      .7  214.06    1.01
  219.82    2.25  235.36    2.14  253.53    2.38  269.09    2.36  318.43    3.15
  329.71    4.21  351.95       5
#Mann= 3 , 0 , 0
       0    .045       0  182.41    .035       0  214.06    .045       0
#XS Ineff= 2 , 0
       0   135.9       5               0
Permanent Ineff=
       F       F
Bank Sta=182.41,214.06
XS Rating Curve= 0 ,0
Exp/Cntr=0.3,0.1

Type RM Length L Ch R = 1 ,425.41  ,33.23,23.41,23.54
Node Photo=..\..\..\Corner Brook\Windshield Survey\CB photos\P1000632.JPG
XS GIS Cut Line= 6
      344912.125       5424006.5      344941.527     5424014.313
      344951.749     5424040.729      345053.649     5424047.601
      345212.438     5424119.444      345291.579     5424095.917
#Sta/Elev= 21
       0       5   58.39    3.87   80.33    3.52  186.34    2.81  186.98    2.79
   191.3    1.64  194.05     1.4  198.77     1.2  199.32   1.012  200.23      .7
  207.79     .48  222.27     .74  222.95     .99  224.98    1.72   249.2    2.63
  251.93    3.05  259.35    3.16  349.01    2.37  359.22    2.73  379.88    3.26
   419.6       5
#Mann= 3 , 0 , 0
       0    .055       0  199.32    .035       0  222.95    .055       0
Bank Sta=199.32,222.95
XS Rating Curve= 0 ,0
Exp/Cntr=0.3,0.1

Type RM Length L Ch R = 1 ,381.26  ,7.2,7.2,7.2
Node Photo=..\..\..\Corner Brook\Windshield Survey\CB photos\P1000628.JPG
XS GIS Cut Line= 6
      344906.781       5424015.5      344934.904     5424020.931
      344938.538     5424044.632      344979.135     5424077.939
      345210.052     5424152.158       345309.16     5424121.075
#Sta/Elev= 29
       0       5   52.62    4.17   96.34    2.81  101.04    2.71  102.31    2.73
  189.03    2.85  197.87    2.83  199.63    2.75  205.53     1.4  207.13    1.32
   207.5    1.25  208.28    1.09  209.47      .9  226.38     .79  229.06     .92
  230.32    1.46   231.1    1.79  235.72    2.22  237.03    2.56  237.63    2.59
  237.64    2.59  280.68    3.21   315.1     2.9  344.56    2.64  354.82     2.7
  365.44    2.86  422.65     2.8  425.91    3.63  451.71       5
#Mann= 3 , 0 , 0
       0    .055       0   207.5    .035       0  230.32    .055       0
#XS Ineff= 2 , 0
   52.62  208.28    2.84  228.98   52.62    2.64
Permanent Ineff=
       F       F
Bank Sta=207.5,230.32
XS Rating Curve= 0 ,0
Exp/Cntr=0.5,0.3

Type RM Length L Ch R = 3 ,380     ,,,
Node Photo=..\..\..\Corner Brook\Windshield Survey\CB photos\P1000626.JPG
BEGIN DESCRIPTION:
Corner Brook Pulp & Paper #3 - Foot Bridge (Structure #2104)
END DESCRIPTION:
Bridge Culvert--1,0,-1,-1, 0
Deck Dist Width WeirC Skew NumUp NumDn MinLoCord MaxHiCord MaxSubmerge Is_Ogee
1.3,4,1.67,0, 6, 6, 2.64, , 0.98, 0, 0,0,,
  189.03  208.28  208.29  228.97  228.98  258.65
    2.84    2.84    2.84    2.84    2.84    2.84
      .9      .9    1.95    1.95      .9      .9
  178.22  197.47  197.48  218.16  218.17  247.84
    2.84    2.84    2.84    2.84    2.84    2.84
      .9      .9    1.95    1.95      .9      .9
BR Coef=-1 , 0 , 0 ,, 0 ,,,0.8,-1,,0,
WSPro=,,,, 1 ,,,, 0 ,,,, 0 ,,,,-1 ,-1 ,-1 , 0 , 0 , 0 , 0 , 0
BC Design=,, 0 ,, 0 ,,,,,,
BC Use User HTab Curves=0
BC User HTab FreeFlow(D)= 0

Type RM Length L Ch R = 1 ,375.14  ,22.33,22.25,22.11
Node Photo=..\..\..\Corner Brook\Windshield Survey\CB photos\P1000623.JPG
XS GIS Cut Line= 6
       344904.25       5424018.5      344926.692     5424022.519
      344929.243     5424041.353      344961.126     5424079.461
      345210.563     5424161.925      345313.322     5424129.032
#Sta/Elev= 23
       0       5   41.81    4.17   90.23    2.71  187.06    2.83  188.82    2.75
  194.72     1.4  196.32    1.32  197.94   1.015  198.66      .9  215.57     .79
  218.25     .92  218.48   1.019  220.29    1.79  224.91    2.22  226.22    2.56
  226.82    2.59  269.87    3.21  333.75    2.64  354.63    2.86  411.84     2.8
  416.13    2.52  438.65    3.63  462.52       5
#Mann= 3 , 0 , 0
       0    .055       0  197.94    .035       0  218.48    .055       0
#XS Ineff= 2 , 0
   41.81  197.47    2.35  218.17   41.81    2.35
Permanent Ineff=
       F       F
Bank Sta=197.94,218.48
XS Rating Curve= 0 ,0
Exp/Cntr=0.5,0.3

Type RM Length L Ch R = 1 ,352.89  ,29.06,28.77,28.44
Node Photo=..\..\..\..\Corner Brook\Windshield Survey\CB photos\P1000622.JPG
BEGIN DESCRIPTION:
Grade change in stream
END DESCRIPTION:
XS GIS Cut Line= 5
      344892.938       5424029.5      344899.236      5424060.72
      344968.628     5424104.451      345216.814     5424179.417
       345318.23     5424148.638
#Sta/Elev= 27
       0       5   31.85     3.5   45.19    3.05   49.47     3.2   67.71    2.96
   70.52    2.51   72.78    2.59  107.82    2.88  128.46     2.9  179.05    3.15
  181.74    2.88  193.33    2.37  196.94   1.014  197.56     .77  207.57     .68
  226.41      .8  227.35   1.042  230.87    1.95     247    2.79   278.7    3.24
   327.4     2.8  336.24    2.84  373.13    3.29  436.28    3.25  444.82    2.68
  461.33    3.53  479.12       5
#Mann= 3 , 0 , 0
       0    .055       0  196.94    .035       0  227.35    .055       0
Bank Sta=196.94,227.35
XS Rating Curve= 0 ,0
Exp/Cntr=0.3,0.1

Type RM Length L Ch R = 1 ,324.13  ,31.82,31.21,30.62
XS GIS Cut Line= 4
344888.6082763675424061.96929932344962.3762817385424133.18768311
345220.5648803715424209.40411377345308.7117309575424176.29370117
#Sta/Elev= 29
       0     3.8   13.94     3.5   28.59    3.42   34.54    2.23   39.29    2.47
   41.68     2.5  116.89    3.11  152.25    3.14  158.58    3.04  162.62    2.91
  178.94    1.88  182.35     .86  182.56      .8  198.39     .67  211.49     .78
   211.8    .859   212.9    1.14  249.12    3.04  266.15    3.28   291.7    3.05
  303.88    3.04  327.81    3.45  371.74    3.34  444.33    3.59  444.45     3.7
  445.07    3.55  447.87    3.48  464.37     3.5   465.9     3.8
#Mann= 3 , 0 , 0
       0    .055       0  182.35    .035       0   211.8    .055       0
Bank Sta=182.35,211.8
XS Rating Curve= 0 ,0
Exp/Cntr=0.3,0.1

Type RM Length L Ch R = 1 ,292.92  ,27.57,18.3,8.5
XS GIS Cut Line= 6
 344882.333923345424066.41009521344951.7260742195424163.86712646
345107.3892822275424207.59771729345131.3881225595424222.67687988
345275.7416992195424249.74768066345338.8267211915424206.36010742
#Sta/Elev= 30
       0     3.8    2.73     3.5   17.11    3.12   22.75    3.28   27.45    2.12
   27.87    2.15   31.89     3.4   35.37    2.78   46.02    2.44  119.64    2.83
  155.08    3.23  191.69    2.49  194.24    1.96   197.7    1.63  199.44   1.165
  201.12     .65  226.12     .87  231.16    1.08  284.97    3.32  395.93    3.71
  431.43    2.86  456.54    3.12  461.77    3.93  467.28    3.04  472.05    3.07
  473.22    3.99  479.15    2.72  502.95    2.38  509.01    2.56   533.1    3.84
#Mann= 3 , 0 , 0
       0    .055       0  199.44    .035       0  231.16    .055       0
Bank Sta=199.44,231.16
XS Rating Curve= 0 ,0
Exp/Cntr=0.3,0.1

Type RM Length L Ch R = 1 ,274.62  ,7.58,7.62,7.75
Node Photo=..\..\..\..\Corner Brook\Windshield Survey\CB photos\P1000620.JPG
XS GIS Cut Line= 6
344852.3264770515424074.53149414344959.4033203135424200.96429443
345105.0242919925424212.23687744345130.6458740235424224.16027832
345276.4838867195424252.34350586345341.0532836915424208.77050781
#Sta/Elev= 30
       0     3.8    2.37     3.5   13.04    3.04   21.04    1.89   61.28    1.96
   77.66    2.91   92.03    2.38  165.68    2.77  198.09    3.11  225.74    2.63
  240.67    1.97  248.95   1.298  253.11     .96  263.72   1.362  306.36    2.98
   319.1    3.29  452.36    3.81  488.54       3  489.47    2.77  497.08    3.94
  503.06    3.04  503.88    3.71  504.45    4.03  505.06    4.04  506.24    3.49
   510.3    2.68  535.66    2.35  545.66    2.64  562.95    3.54  566.43    3.84
#Mann= 3 , 0 , 0
       0    .055       0  248.95    .035       0  263.72    .055       0
#XS Ineff= 2 , 0
       0  242.99    1.89  269.06       0    1.85
Permanent Ineff=
       F       F
Bank Sta=248.95,263.72
XS Rating Curve= 0 ,0
Exp/Cntr=0.5,0.3

Type RM Length L Ch R = 1 ,245.99  ,31.94,35.1,38.27
XS GIS Cut Line= 5
      344843.574      5424078.28      344954.227     5424218.843
       345109.89     5424250.704      345296.811     5424309.428
      345384.333      5424248.83
#Sta/Elev= 30
       0     3.8     1.2     3.5    7.02     3.1    10.6    2.25   12.67    1.93
   92.75    2.09  103.58    2.67  112.74    2.35  178.89     2.6  221.94       3
  231.03    2.87  240.11    2.48  242.29   1.458  243.38     .95  254.36     .64
  260.54    1.47  263.91    1.92   279.1    1.56  317.69    2.76  329.35     2.9
  330.88    2.27  340.82    3.11  484.25    3.71  514.08    3.65  541.63    2.91
  548.95    2.07  564.92    2.41  627.86    3.03  638.27    3.48  640.16     3.8
#Mann= 3 , 0 , 0
       0    .055       0  242.29    .035       0  260.54    .055       0
Bank Sta=242.29,260.54
XS Rating Curve= 0 ,0
Exp/Cntr=0.3,0.1

Type RM Length L Ch R = 1 ,210.89  ,38.68,35.99,33.1
XS GIS Cut Line= 6
      344842.324     5424080.779      344906.715      5424214.47
      344933.596     5424244.456      345101.138     5424290.061
      345303.688     5424320.673      345404.963     5424265.697
#Sta/Elev= 28
       0       5    4.13       4   10.23    3.55   52.68     3.6  133.57    3.08
  173.47    2.91  189.06    1.57   194.4    1.96  195.79    2.57  229.71    2.39
  237.99    1.92  262.78    1.42  283.86     .68   284.7   1.438  287.41    2.92
  290.45       3  355.75    2.39  360.11    2.72  371.98    3.04  389.61    2.33
  405.78    2.29  414.27    2.58  417.98    2.28  493.81    1.97  541.16    1.94
  545.69    3.13  661.06       4  682.38       5
#Mann= 3 , 0 , 0
       0    .055       0  262.78    .035       0   284.7    .055       0
Bank Sta=262.78,284.7
XS Rating Curve= 0 ,0
Exp/Cntr=0.3,0.1

Type RM Length L Ch R = 1 ,174.77  ,22.25,19.11,16.6
XS GIS Cut Line= 5
      344757.928     5424108.891      344937.972     5424287.562
      345203.663     5424341.913      345311.815     5424347.536
      345414.965     5424275.068
#Sta/Elev= 30
       0       4    8.81    2.09   51.34    3.34  120.15    3.36  218.42    2.84
  224.78    3.06  246.67    3.18  293.16    2.25   303.4    2.19  308.15   1.934
  319.52    1.32  322.52     .69  332.76    1.14  335.93    2.01  339.41    3.03
  346.21    2.31   388.3    2.07  423.29    2.35  428.78    2.84  431.71    2.63
  470.25    2.25  499.77    3.35  518.36    2.21  629.98    1.63  630.35    1.55
  632.66    2.03  635.32    2.41  641.92    3.81  733.15       4   759.2       5
#Mann= 3 , 0 , 0
       0    .055       0  308.15    .035       0  335.93    .055       0
Bank Sta=308.15,335.93
XS Rating Curve= 0 ,0
Exp/Cntr=0.3,0.1

Type RM Length L Ch R = 1 ,155.66  ,6.01,5.58,5.11
Node Photo=..\..\..\Corner Brook\Windshield Survey\CB photos\P1000612.JPG
XS GIS Cut Line= 5
      344662.905     5424187.607      344939.848     5424311.302
      345201.162     5424348.161      345311.815     5424351.909
      345420.591     5424277.567
#Sta/Elev= 30
       0       6    1.54       5    21.8       3   23.57    2.57   36.22    1.75
   88.59     3.3   162.5    3.32  263.15    2.85  276.38     3.3  291.02    3.42
  336.33    2.61  344.93    2.08  355.72    2.16  366.56    1.32  370.92     .64
  372.17   1.483  373.59    2.08  375.16     2.6  382.29    2.15  411.58    2.06
  417.88    2.24  430.26     1.9  443.51    1.89  511.86    2.27  557.05    2.02
  676.56    2.35  781.39       3  803.97       4  808.43       5  809.68       6
#Mann= 3 , 0 , 0
       0    .055       0  355.72    .035       0  373.59    .055       0
#XS Ineff= 2 , 0
       0  355.72    2.08  373.59       0    1.89
Permanent Ineff=
       F       F
Bank Sta=355.72,373.59
XS Rating Curve= 0 ,0
Exp/Cntr=0.4,0.2

Type RM Length L Ch R = 1 ,150.09  ,8.19,21.03,33.59
Node Photo=..\..\..\Corner Brook\Windshield Survey\CB photos\P1000610.JPG
XS GIS Cut Line= 5
      344657.904     5424193.854      344946.099     5424318.174
      345198.037     5424350.659       345313.69     5424356.907
      345423.717     5424282.565
#Sta/Elev= 30
       0       6     1.1       5   21.03       4   86.09    3.28  161.96     3.3
  221.01    2.92  262.85    2.86   278.4    3.38  290.49    3.49  325.33    2.88
  338.75    2.06  354.83    2.09  363.56    1.48  368.61     .55  370.41    1.24
  378.07   2.077  380.93    2.39  401.95    2.18   411.9    2.43  429.89    1.93
  505.42    2.23  554.96    2.01  643.15    2.29  667.43       2  706.63       2
  789.62       3  798.21       4  814.33       5  815.24       6   816.5       7
#Mann= 3 , 0 , 0
       0    .055       0  354.83    .035       0  378.07    .055       0
#XS Ineff= 2 , 0
       0  354.83    2.06  378.07       0    1.91
Permanent Ineff=
       F       F
Bank Sta=354.83,378.07
XS Rating Curve= 0 ,0
Exp/Cntr=0.4,0.2

Type RM Length L Ch R = 1 ,129.05  ,48.12,48.32,47.32
XS GIS Cut Line= 5
      344650.402     5424196.353      344946.099     5424325.046
      345052.376     5424371.275       345314.94     5424361.904
      345427.468     5424287.562
#Sta/Elev= 30
       0       8    1.08       7     2.9       6    5.57       5   24.33       4
   38.08       3   83.26    3.21  285.42     2.9  296.64    3.26  301.83    5.83
   311.2    6.57   320.3    2.78  329.09    2.55  355.45    1.26  369.46    1.08
  380.53      .4  381.21   1.234  384.24    2.58  390.04    2.43  410.86     2.7
  437.31    1.97   521.5    2.21  559.94       2  647.23    2.26  685.77       2
  726.23       2  809.44       3  833.62       5  835.52       7  835.98       8
#Mann= 3 , 0 , 0
       0    .055       0  355.45    .035       0  381.21    .055       0
Bank Sta=355.45,381.21
XS Rating Curve= 0 ,0
Exp/Cntr=0.3,0.1

Type RM Length L Ch R = 1 ,80.73   ,61.44,56.94,50.51
XS GIS Cut Line= 6
      344609.509     5424239.208      344674.667     5424295.925
      345003.964     5424402.357      345082.434     5424375.749
      345317.145     5424365.246      345430.647     5424289.623
#Sta/Elev= 30
       0       6   15.38       5   86.42       4   90.25    3.18  261.49    2.93
  280.63    3.02  287.18    5.06   309.4    4.47  314.06    7.16  323.23    7.48
  327.16    7.23   338.1    2.09  354.99    1.69  358.19    3.11  363.51     3.6
  369.86    1.03  376.11     .81  378.91      .2  403.76     .85  410.81    3.72
  481.14    5.45  499.25    5.28  505.82       3  518.84    2.25     539    3.04
  608.87    1.76  777.28       2  860.94       3  884.12       5  887.98       8
#Mann= 3 , 0 , 0
       0    .055       0  376.11    .035       0  403.76    .055       0
Bank Sta=376.11,403.76
XS Rating Curve= 0 ,0
Exp/Cntr=0.3,0.1

Type RM Length L Ch R = 1 ,23.81   ,26,23.8,24.26
XS GIS Cut Line= 6
      344581.484     5424256.713      344642.438     5424323.933
      344875.748     5424417.761      345020.779     5424453.472
      345319.247     5424369.447       345433.45     5424293.124
#Sta/Elev= 30
       0       7   13.67       5  132.18    2.94  278.01     2.2   291.5    2.88
  326.26    2.63  331.69    3.57  334.97    6.29  347.76    8.44  373.57    8.84
  378.62    8.65  384.84    6.41  391.86    1.93  394.97    1.04  404.26     .32
  430.52     .88  431.89    1.65  435.95    3.26  449.49    4.52  499.58    3.15
  502.73    1.72  508.67    3.42  535.57    5.05  556.33    3.57   616.2    3.12
  627.38    1.62  913.66       3  923.64       5  937.79       6  939.51       7
#Mann= 3 , 0 , 0
       0    .055       0  391.86    .035       0  431.89    .055       0
Bank Sta=391.86,431.89
XS Rating Curve= 0 ,0
Exp/Cntr=0.3,0.1

--- Corner_Brook2.g03 (geometry) ---

Geom Title=CB_with_below_waterline_gates
Program Version=4.10
BEGIN GEOM DESCRIPTION:
Created based on a TIN with 1 z tolerance
END GEOM DESCRIPTION:

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
River Reach=BellsB          ,TR001

Type RM Length L Ch R = 1 ,178.13  ,18.25,18.27,18.06
XS GIS Cut Line= 6
344234.4996948245422720.95068359344238.9260864265422731.27270508
344238.0407104495422749.41009521344253.2380981455422758.25750732
344279.2062988285422758.69989014344288.9442749025422755.16088867
#Sta/Elev= 29
       0   100.6    1.07  100.17    1.36   100.1    3.95   99.29    6.84   98.69
   11.23   98.43   26.64   97.18   26.75   97.17   29.39   97.06   29.64   97.06
    33.3   95.27   34.92    94.8    37.4   93.66   38.11   93.33   39.46   93.14
   39.72   92.91   40.89  93.708   43.36   94.97   44.56    95.4   46.98   96.42
    48.3   96.87   49.69   96.98   50.19   97.07   66.89      98   72.95   99.37
    79.9  100.72   80.71  100.84   82.12  100.98   83.31  101.11
#Mann= 3 , 0 , 0
       0    .055       0    37.4    .035       0   40.89    .055       0
Bank Sta=37.4,40.89
XS Rating Curve= 0 ,0
Exp/Cntr=0.3,0.1

Type RM Length L Ch R = 1 ,159.86  ,19.69,20.32,20.7
XS GIS Cut Line= 2
344199.8156738285422748.48608398344269.362304688 5422788.0244751
#Sta/Elev= 25
       0  100.72    5.48   98.62    7.71   97.22   12.75   96.95   16.31   96.67
   22.63   96.54   26.89   96.37   32.21   96.16   32.29   96.14   33.23   95.54
   38.95   92.89      39   92.86   39.61   92.56   40.09   92.15   40.73   92.43
      41   92.46   42.58  92.644   44.18   92.83   45.24   93.38   51.06   96.33
   59.79   96.63    70.5   96.86   73.81   96.97   79.98   98.32      80   98.32
#Mann= 3 , 0 , 0
       0    .055       0   39.61    .035       0   42.58    .055       0
Bank Sta=39.61,42.58
XS Rating Curve= 0 ,0
Exp/Cntr=0.3,0.1

Type RM Length L Ch R = 1 ,139.54  ,49.06,48.13,33.83
Node Photo=..\..\..\..\Corner Brook\Windshield Survey\CB photos\P1000709.JPG
XS GIS Cut Line= 5
       344187.04     5422775.179      344200.338      5422782.01
      344217.269     5422780.434      344217.269     5422780.434
      344255.016     5422806.982
#Sta/Elev= 30
       0     100     1.7      99    3.45      98    5.35      97    7.53      96
   10.51      95   14.95      96   24.47      96   26.94   96.28   32.46   96.28
   33.74      96   35.57      95   36.96      94   38.56      93   38.84   93.02
  38.845   92.11   38.85   91.14   38.92   91.14   39.81   91.14   40.26   91.13
    41.3   91.13   41.31   92.11   42.23    92.2   43.18      93   46.09      94
   47.56      95   49.89      96   52.35      97   60.24   97.09    78.1   97.09
#Mann= 3 , 0 , 0
       0    .055       0  38.845    .035       0   41.31    .055       0
#XS Ineff= 2 , 0
       0   38.92   96.28   41.32       0   96.78
Permanent Ineff=
       F       F
Bank Sta=38.845,41.31
XS Rating Curve= 0 ,0
Exp/Cntr=0.5,0.3

Type RM Length L Ch R = 2 ,100     ,,,
Node Photo=..\..\..\..\Corner Brook\Windshield Survey\CB photos\P1000708.JPG
BEGIN DESCRIPTION:
O'Connell Drive/Mount Batten Road (Structure #2130)
END DESCRIPTION:
Bridge Culvert--1,0,-1,-1, 0
Deck Dist Width WeirC Skew NumUp NumDn MinLoCord MaxHiCord MaxSubmerge Is_Ogee
12,19.2,1.67,0, 7, 8, 95, , 0.98, 0, 0.73,0.57,,
       0    5.44    24.2   31.78   37.33   52.04   63.15
   95.92   95.85   96.78      97   97.05      97   97.09
                                                        
       0   19.48   28.32   36.51   40.19   45.24   49.91   66.38
      97   95.92   95.85      96      96   95.71   95.42      97
                                                                
BR Coef=-1 , 0 , 0 ,, 0 ,,,0.8,-1,,0,
WSPro=,,,, 1 ,,,, 0 ,,,, 0 ,,,,-1 ,-1 ,-1 , 0 , 0 , 0 , 0 , 0
Culvert=1,2.4,,44.2,0.03,0.7,1,2,2,91.13,40.12,89.49,40.27,Culvert #1  , 0 ,1.4
Culvert Bottom n=0.03
BC Design=,, 0 ,, 0 ,,,,,,
BC Use User HTab Curves=0
BC User HTab FreeFlow(D)= 0

Type RM Length L Ch R = 1 ,91.42   ,3.23,3.25,0.95
Node Photo=..\..\..\..\Corner Brook\Windshield Survey\CB photos\P1000713.JPG
XS GIS Cut Line= 6
344176.3275146485422793.74768066344187.5899047855422816.60327148
344192.6146850595422823.52929688344201.1046752935422826.99230957
344212.5405273445422816.77648926344218.2583007815422811.40887451
#Sta/Elev= 19
       0      97   27.82      96    29.8      95   31.53      94   33.34      93
    36.2      92   38.17   91.55   38.37      90   39.17  89.759   40.06   89.49
   40.82   89.49   41.03   89.49   41.29  89.933   41.94   91.04   43.13      91
   46.01      92   49.33      93   52.76      94   66.38      96
#Mann= 3 , 0 , 0
       0    .055       0   38.37    .035       0   41.29    .055       0
#XS Ineff= 2 , 0
       0   39.07   93.65   41.47       0   93.65
Permanent Ineff=
       F       F
Bank Sta=38.37,41.29
XS Rating Curve= 0 ,0
Exp/Cntr=0.5,0.3

Type RM Length L Ch R = 1 ,88.17   ,2.5,4.05,10.03
XS GIS Cut Line= 6
344174.2482910165422796.34509277344185.5106811525422819.20068359
344190.5355224615422826.12652588344199.0255126955422829.58947754
344210.4613037115422819.37371826344216.1790771485422814.00610352
#Sta/Elev= 24
       0   97.07   25.47   96.22   25.48   96.21   34.04   92.08   34.66   91.89
   34.86   91.86   35.62   91.59   36.82   90.72   39.14   89.63   39.42   89.47
   40.45  88.864   40.78   88.47   41.92   88.75   43.21   88.84   44.37    89.1
   47.56   91.21    56.5   94.19   57.23   94.44   57.28   94.45   57.55   94.52
   58.54   94.81   61.75   95.78   63.05   95.86   66.38   95.95
#Mann= 3 , 0 , 0
       0    .055       0   40.45    .035       0   43.21    .055       0
Bank Sta=40.45,43.21
XS Rating Curve= 0 ,0
Exp/Cntr=0.3,0.1

Type RM Length L Ch R = 1 ,84.12   ,3.03,4.98,8.8
XS GIS Cut Line= 6
344172.6889038095422796.34509277344187.4166870125422824.04870605
344193.3076782235422831.49407959344199.372070313 5422834.0914917
344213.0603027345422825.26068115344222.7633056645422817.64227295
#Sta/Elev= 24
       0   97.12   26.05   96.23   31.38   93.56   35.51   91.59   35.77   91.44
    36.2   91.36   36.38   91.33   37.44   91.06    39.2   90.27   40.87   89.28
   41.55   88.88   42.87  88.102   43.28   87.66   44.32   87.93   47.47   88.14
   51.66   89.03   52.72   89.72   55.22   90.47   61.86   94.27   63.76   94.37
   68.59   94.62    71.2   95.37   71.88   95.41   76.09   95.49
#Mann= 3 , 0 , 0
       0    .055       0   42.87    .035       0   47.47    .055       0
Bank Sta=42.87,47.47
XS Rating Curve= 0 ,0
Exp/Cntr=0.3,0.1

Type RM Length L Ch R = 1 ,79.14   ,5.7,6.39,8.69
XS GIS Cut Line= 6
344172.5156860355422797.38391113344184.6442871095422820.23950195
344189.4959106455422830.80151367344192.6146850595422836.86169434
 344198.505676275422838.07373047344222.416687012 5422829.4163208
#Sta/Elev= 26
       0    97.1     .01    97.1   25.05   96.24   25.87   95.83    32.9   92.27
   34.18   91.47    37.5   90.71   37.59   90.69   38.88    90.5   39.24   90.38
   43.48   87.68   44.31   87.19   44.77    86.9   45.02   86.74   46.21   86.53
   47.05   86.79   47.47   86.88   47.98   86.97   50.33   87.37   51.24   87.61
   57.01   88.77   60.07   90.49   61.37   91.24   66.36   94.17   72.64   94.49
   75.76   94.63
#Mann= 3 , 0 , 0
       0    .055       0   44.77    .035       0   47.98    .055       0
Bank Sta=44.77,47.98
XS Rating Curve= 0 ,0
Exp/Cntr=0.3,0.1

Type RM Length L Ch R = 1 ,72.74   ,2.71,4.99,10
XS GIS Cut Line= 6
344171.8225097665422799.11547852344184.1245117195422820.93212891
344188.6295166025422839.97851563344193.3076782235422843.78771973
344216.6989135745422842.22930908344227.2681274415422834.95709229
#Sta/Elev= 18
       0   97.04   23.65   96.26   30.25    92.9   32.42   91.49   38.36    90.1
   45.04   88.05   47.79  86.196   48.14   85.76   52.44   86.18   56.09   86.69
   57.64   86.63   61.27   87.56   64.46   89.61   70.49   93.88   71.28   93.99
   75.63   94.03   84.82   94.49   86.94   94.73
#Mann= 3 , 0 , 0
       0    .055       0   47.79    .035       0   52.44    .055       0
Bank Sta=47.79,52.44
XS Rating Curve= 0 ,0
Exp/Cntr=0.3,0.1

Type RM Length L Ch R = 1 ,67.75   ,2.94,3.71,5.31
XS GIS Cut Line= 5
344170.9561157235422800.32751465344182.3919067385422821.62469482
344188.1096801765422845.86547852344201.4512939455422856.25427246
344215.1395263675422858.85168457
#Sta/Elev= 27
       0   96.98    3.31   96.96   22.52    96.3   24.17   95.47   28.09   93.47
   31.11   91.51   35.87    90.4   36.19   90.28    38.9   89.55   48.29   86.66
   49.08    86.4   49.29   86.34   50.28   85.67   50.92   85.04   55.32   85.35
   55.94   85.37   56.12   85.36   58.28   85.46   59.78   87.57   60.83   88.77
   62.39   90.67   62.61      91   65.25    92.8   65.99   92.96   66.38   93.03
   72.89    93.3   79.92   93.41
#Mann= 3 , 0 , 0
       0    .055       0   50.28    .035       0   55.32    .055       0
Bank Sta=50.28,55.32
XS Rating Curve= 0 ,0
Exp/Cntr=0.3,0.1

Type RM Length L Ch R = 1 ,64.04   ,3.68,3.35,4.35
XS GIS Cut Line= 5
344169.7432861335422800.50048828344180.4859008795422821.27832031
344182.5651245125422830.97467041344185.8572998055422847.59692383
344200.5848999025422866.29711914
#Sta/Elev= 26
       0   96.95    6.05    96.9   22.56   96.34   23.39   95.92   27.06   94.05
   30.93   91.53   33.31   90.97    34.4   90.72   34.92   90.53   39.51   89.28
   50.25   85.97   51.74   85.58   53.17    85.2   53.39   85.13   54.06    84.7
   56.42   84.47   57.07   84.72   59.16   85.17   62.57   89.71   62.64   89.81
   62.73   89.92   63.32   90.84   64.14   92.12    64.2   92.13   66.17   92.54
   74.06   92.49
#Mann= 3 , 0 , 0
       0    .055       0   53.39    .035       0   59.16    .055       0
Bank Sta=53.39,59.16
XS Rating Curve= 0 ,0
Exp/Cntr=0.3,0.1

Type RM Length L Ch R = 1 ,60.69   ,4.56,3.94,4.31
XS GIS Cut Line= 5
344164.1987304695422804.13671875344179.4462890635422833.39868164
 344182.738281255422847.25067139344187.9362792975422857.12011719
344197.6392822275422868.20172119
#Sta/Elev= 27
       0   96.71   18.01   96.56   20.34   96.48   21.09    96.1    28.4   91.58
   29.05   91.43   30.29   91.03      33   90.35   38.48   88.87   47.23   86.18
   50.88   85.13   52.04    84.8   53.43   84.14   55.58   84.69   55.79   84.72
   56.44   84.85   58.39   85.29   58.71   85.36   59.59   86.31   60.14   86.85
   61.16   88.51   63.18   91.86   64.13   91.99   64.96   92.34   65.02   92.35
   66.87   92.33   73.12   92.32
#Mann= 3 , 0 , 0
       0    .055       0   50.88    .035       0   55.58    .055       0
Bank Sta=50.88,55.58
XS Rating Curve= 0 ,0
Exp/Cntr=0.3,0.1

Type RM Length L Ch R = 1 ,56.76   ,7.72,5.83,4.41
XS GIS Cut Line= 4
344158.3076782235422827.16552734 344178.579895025422847.07751465
344186.7235107425422864.21929932344193.4810791025422870.10632324
#Sta/Elev= 23
       0   96.48    5.04    96.4    8.11   93.83   11.37   92.34   15.68   89.62
   18.36   88.67   21.86   87.95   28.42   86.38   31.19   85.57   33.47   84.81
   35.37   83.97   38.73   84.71   40.25   84.96   41.38   85.13   42.15   87.01
   43.35    87.9   44.82   90.58   44.99   90.62   46.16   91.45   47.39   91.98
   47.99   92.23   48.26   92.31   56.36    92.2
#Mann= 3 , 0 , 0
       0    .055       0   33.47    .035       0   38.73    .055       0
Bank Sta=33.47,38.73
XS Rating Curve= 0 ,0
Exp/Cntr=0.3,0.1

Type RM Length L Ch R = 1 ,50.93   ,7.48,7.07,7.18
XS GIS Cut Line= 3
344154.1492919925422830.97467041344182.045288086 5422862.4876709
344192.0949096685422870.62567139
#Sta/Elev= 27
       0   96.43    4.55   96.35    5.62   95.45    8.95   93.95    9.45   93.86
   12.53   91.66   14.82   90.06   19.75   87.21   20.66   86.81   21.68   86.49
   27.38   84.93   28.89   84.55   30.17  84.189   30.91   83.98   31.27   83.68
   31.63   83.94   36.01   84.58   38.61   84.95   40.23   88.54   41.68   90.29
   42.09   90.24   42.78   90.17   44.72   91.09   45.71    91.8    46.7   92.19
   47.04    92.3   55.02   92.19
#Mann= 3 , 0 , 0
       0    .055       0   30.17    .035       0   36.01    .055       0
Bank Sta=30.17,36.01
XS Rating Curve= 0 ,0
Exp/Cntr=0.3,0.1

Type RM Length L Ch R = 1 ,43.86   ,6.35,6.86,7.11
XS GIS Cut Line= 3
344148.4312744145422837.38128662344180.3126831055422869.93310547
344188.4562988285422875.99328613
#Sta/Elev= 20
       0   96.52    4.55   95.97   12.51   89.96   12.71   89.84   14.08   88.75
   14.25   88.65   14.38   88.55   26.94  83.804   27.48    83.6   27.99   83.34
   28.14   83.59   33.56   84.03   35.67    84.2   39.14   88.33   41.47   89.96
   45.36    92.2   45.56    92.2   47.15   92.23   50.35   92.17   55.71    92.1
#Mann= 3 , 0 , 0
       0    .055       0   26.94    .035       0   33.56    .055       0
Bank Sta=26.94,33.56
XS Rating Curve= 0 ,0
Exp/Cntr=0.3,0.1

Type RM Length L Ch R = 1 ,37.01   ,27.23,24.86,22.79
XS GIS Cut Line= 3
344145.4793090825422841.12591553344173.7730712895422874.27587891
 344184.958923345422878.58673096
#Sta/Elev= 19
       0   96.14    4.25   95.62    8.93   92.07   10.99   90.63   13.32   90.19
   13.73   89.97   18.66   86.27    25.7   83.58   27.09   83.43   29.82   82.98
   30.72   83.51   32.12   83.62    33.8   83.75   35.14   85.35   43.58   91.17
   44.18   91.57   45.06   92.04   50.26   92.15   55.57   92.07
#Mann= 3 , 0 , 0
       0    .055       0   27.09    .035       0   32.12    .055       0
Bank Sta=27.09,32.12
XS Rating Curve= 0 ,0
Exp/Cntr=0.3,0.1

Type RM Length L Ch R = 1 ,12.14   ,4.7,12.15,6.96
XS GIS Cut Line= 6
344139.0648803715422843.84472656344136.9857177735422848.86608887
344142.5302734385422874.31890869344145.1292724615422880.89849854
344157.6044921885422887.30487061344184.6342773445422879.51330566
#Sta/Elev= 29
       0    96.1    5.43   95.84    5.48   95.84   13.26   92.56   14.37    91.9
   15.84   91.54   17.28   91.32   21.12   90.73   25.12   89.93   29.84   88.78
   31.48   87.72   31.88   87.46   34.77   85.25   38.56   82.95   39.11  82.606
   39.52   82.15    40.9   82.42   45.09   82.63   46.48   82.65   47.95   82.68
   50.31   84.26   52.58   85.06   57.87   87.62    58.5   87.85   63.47   89.97
   63.73   90.05   70.56   91.99   74.61    92.1   80.71   92.06
#Mann= 3 , 0 , 0
       0    .055       0   39.11    .035       0   45.09    .055       0
Bank Sta=39.11,45.09
XS Rating Curve= 0 ,0
Exp/Cntr=0.3,0.1

River Reach=BellsB          ,M002

Type RM Length L Ch R = 1 ,5166.11 ,15.85,16.88,18.06
XS GIS Cut Line= 2
342277.9199218755421174.32928467342246.3927001955421094.99212646
#Sta/Elev= 21
       0  194.87    4.87  193.53    5.46  193.51   16.24  192.65    24.2  192.33
   30.49  193.13   33.24   192.5   35.69  191.76   36.61  191.67   44.35  191.12
   46.35  190.98   47.49  190.79   48.76 191.067   51.01  191.38   57.79  192.95
   61.01  193.34   61.28  193.35   67.04  193.71   80.92  194.96   81.94   195.1
   85.37  195.66
#Mann= 3 , 0 , 0
       0    .065       0   46.35     .04       0   48.76    .065       0
Bank Sta=46.35,48.76
XS Rating Curve= 0 ,0
Exp/Cntr=0.3,0.1

Type RM Length L Ch R = 1 ,5149.23 ,31.28,31.78,26.26
XS GIS Cut Line= 3
342284.6198730475421175.58990479342286.6940917975421159.00872803
 342266.990295415421094.41052246
#Sta/Elev= 21
       0  195.47    3.49  193.81    3.84   193.8   16.71   193.3   25.53  192.92
   29.75  192.59   30.83  192.56   32.16  192.51   37.45  191.29   43.45 190.867
   46.25  190.57   47.35  190.89   49.51  191.32   51.06  191.63   58.15  193.33
   58.71  193.48   63.94  193.76   64.25  193.76   64.35  193.77   65.97  193.87
   84.25  195.04
#Mann= 3 , 0 , 0
       0    .065       0   43.45     .04       0   47.35    .065       0
Bank Sta=43.45,47.35
XS Rating Curve= 0 ,0
Exp/Cntr=0.3,0.1

Type RM Length L Ch R = 1 ,5117.45 ,19.84,26.6,30.57
XS GIS Cut Line= 3
342310.9426879885421195.21392822342324.6160888675421164.53149414
342286.500915527  5421097.578125
#Sta/Elev= 22
       0  194.13   25.55  193.85   33.59   194.1   38.54  194.16   41.05  193.98
   50.37  192.64   55.56  192.13   57.66   191.8   62.74 190.128    63.1  189.91
   64.68 190.056   69.63   190.2   71.63  190.26   72.67  190.29   81.52  191.19
   85.37  192.19   88.35  192.79    88.8  192.82    89.2  192.89   90.21  192.41
   92.38  192.75  110.63  193.96
#Mann= 3 , 0 , 0
       0    .065       0   62.74     .04       0   64.68    .065       0
Bank Sta=62.74,64.68
XS Rating Curve= 0 ,0
Exp/Cntr=0.3,0.1

Type RM Length L Ch R = 1 ,5090.85 ,11.72,23.38,30.25
XS GIS Cut Line= 5
342312.2744750985421195.62567139342333.3610839845421161.42669678
342330.595703125 5421119.2824707 342333.706909185421078.17468262
342337.5092773445421065.39331055
#Sta/Elev= 27
       0   194.1   22.87  193.79   40.18  194.32   41.65  194.36   47.43  193.94
   53.42  193.07   56.52  191.95   68.58  190.24   69.99     190   71.67  189.62
   72.07   189.9   76.71  192.03   78.35  192.54   79.25  193.21   79.73  193.31
   80.68  193.35   82.41  193.39  108.53  193.95  112.89  194.13  118.19  195.39
  119.36  195.97  120.17  196.21  123.64  196.42  123.87  196.44  125.17   196.4
  133.58  197.27  136.97  197.94
#Mann= 3 , 0 , 0
       0    .065       0   69.99     .04       0   72.07    .065       0
#XS Ineff= 2 , 0
       0   41.65  194.36               0
Permanent Ineff=
       F       F
Bank Sta=69.99,72.07
XS Rating Curve= 0 ,0
Exp/Cntr=0.3,0.1

Type RM Length L Ch R = 1 ,5067.47 ,48.56,49.69,45.53
XS GIS Cut Line= 4
342313.2647094735421195.98748779342339.321716309 5421161.1796875
342343.9644775395421135.16009521342390.2396850595421118.28967285
#Sta/Elev= 28
       0  194.08   21.43  193.76   43.48  194.43   44.88  194.47   53.25  193.91
   54.99  193.68   55.73  193.41   57.98  193.15   59.14  192.97      63  192.04
   69.91  190.81   71.59  190.71   74.24  189.32   77.36   189.3   78.38  189.18
   79.36   189.3   81.97  189.31   83.39  190.15   84.24   190.4   84.95  190.83
   87.31  191.88   89.04  192.69   95.49  192.94   96.14  192.88   99.25  192.84
  105.49  192.56  109.43  193.46  119.17  194.07
#Mann= 3 , 0 , 0
       0    .065       0   77.36     .04       0   79.36    .065       0
#XS Ineff= 2 , 0
       0   44.88  194.47               0
Permanent Ineff=
       F       F
Bank Sta=77.36,79.36
XS Rating Curve= 0 ,0
Exp/Cntr=0.3,0.1

Type RM Length L Ch R = 1 ,5017.78 ,49.08,50.21,50
XS GIS Cut Line= 3
 342317.392517095421198.30810547342365.3787231455421178.71252441
342418.3422851565421133.77050781
#Sta/Elev= 24
       0  194.11   18.61  194.11   39.21  194.11   51.83  194.09   63.38  194.18
   63.57  194.08   64.28  193.73    71.6  189.27   74.56  188.62   75.65  188.42
   76.84  188.12   77.65   188.3   83.16  188.89   84.81  189.71   86.95  190.68
   87.54  191.09   87.92  191.33   89.35   192.3   92.31  193.42   95.07  194.66
   97.02  194.78   106.3  195.04  111.18  195.38  121.29  195.93
#Mann= 3 , 0 , 0
       0    .065       0   75.65     .04       0   77.65    .065       0
#XS Ineff= 2 , 0
       0   63.38  194.18               0
Permanent Ineff=
       F       F
Bank Sta=75.65,77.65
XS Rating Curve= 0 ,0
Exp/Cntr=0.3,0.1

Type RM Length L Ch R = 1 ,4967.57 ,45.92,50.1,48.87
XS GIS Cut Line= 6
342356.3491210945421232.34228516342385.2438964845421220.99768066
342427.9514770515421189.73413086342426.5952758795421173.13287354
 342416.976684575421160.14831543342421.3626708985421134.88031006
#Sta/Elev= 28
       0  194.49   24.59  193.83    25.1  193.66   27.15  193.71   31.04  193.56
   40.92  193.16   47.29  189.87   52.49   187.2   53.57  186.55   54.49  186.78
   55.45  186.91   58.38  187.51   64.24  191.22   65.84  191.81   66.05   191.9
   72.02  192.65   83.97  192.17   87.42  192.03   91.08   192.8  100.63  193.39
  108.69  193.98  113.27  194.54  116.79  194.68  129.77  195.28   132.6   195.5
  137.39  195.53   141.9  195.98  142.43     196
#Mann= 3 , 0 , 0
       0    .065       0   52.49     .04       0   54.49    .065       0
Bank Sta=52.49,54.49
XS Rating Curve= 0 ,0
Exp/Cntr=0.3,0.1

Type RM Length L Ch R = 1 ,4917.46 ,19.17,44.16,54.69
XS GIS Cut Line= 6
342357.8818969735421262.62231445 342432.634704595421247.08508301
342461.317871094 5421216.9163208342469.8649291995421203.72247314
342491.2780761725421192.89349365342526.8798828135421141.00531006
#Sta/Elev= 23
       0  194.19   40.11  193.67   49.66  191.92   55.26  188.11   56.48  187.75
   67.37  186.39   76.23  188.14   76.67  188.12   77.24  187.96   82.26  185.81
   83.82  185.69   85.67  185.87   91.56  185.89   92.94  186.53   99.38  190.01
  148.09  189.96  151.23  190.19  162.06  190.26  169.52  190.43  193.67  192.13
  210.51  194.03  213.95  194.31  220.62   194.6
#Mann= 3 , 0 , 0
       0    .065       0   82.26     .04       0   85.67    .065       0
Bank Sta=82.26,85.67
XS Rating Curve= 0 ,0
Exp/Cntr=0.3,0.1

Type RM Length L Ch R = 1 ,4873.31 ,21.46,19.89,10.45
XS GIS Cut Line= 4
342358.6434936525421270.36907959342438.6124877935421267.15551758
342445.2736816415421278.15710449342491.5441284185421265.21850586
#Sta/Elev= 30
       0  194.11    35.5  193.61   37.89  193.54   43.94  193.08   46.92   192.6
   47.42  192.44   55.33  187.31   55.68  187.19   66.45  187.35   73.94  186.69
   76.96  186.27   80.03  186.81   81.22  186.78   85.82  184.88   86.44  184.61
   87.82   185.2   89.97  185.87   94.68  187.08  101.43  187.22   105.2  188.17
  106.36  188.63  107.34  188.82  114.35  191.27  117.64  191.51  120.79  190.67
   123.7  190.95  126.56  190.92  132.13  193.27  134.49  193.35  140.94     194
#Mann= 3 , 0 , 0
       0    .065       0   85.82     .04       0   87.82    .065       0
Bank Sta=85.82,87.82
XS Rating Curve= 0 ,0
Exp/Cntr=0.3,0.1

Type RM Length L Ch R = 1 ,4785.76 ,29.07,29.11,29.57
XS GIS Cut Line= 4
342381.8477172855421362.48071289342405.0465087895421351.04650879
 342451.236511235421353.20410156342487.4505004885421330.52331543
#Sta/Elev= 23
       0  191.79   11.47   190.1   11.65  190.08   11.78  190.07   11.92  190.05
   13.91  189.77   25.86  188.34   27.17  188.12    53.6  181.71    54.2 181.581
   54.58  181.35    55.1  181.52    57.1   181.6   57.25   181.6   58.13  181.96
   61.53  184.66   62.79   185.1   62.85  185.12   66.84  185.01   70.98  185.32
    72.1  185.38   89.47  186.85  114.83  188.92
#Mann= 3 , 0 , 0
       0    .057       0    54.2     .04       0    57.1    .057       0
Bank Sta=54.2,57.1
XS Rating Curve= 0 ,0
Exp/Cntr=0.3,0.1

Type RM Length L Ch R = 1 ,4756.65 ,30.95,29.11,26.42
XS GIS Cut Line= 3
342393.0432739265421378.32452393342446.4367065435421382.54150391
342470.5885009775421367.50811768
#Sta/Elev= 19
       0  188.53    9.27  187.54   18.62  185.87   20.92  185.56   28.55  181.82
   30.15  181.09   33.92  180.71   37.43 180.352   38.72  180.12      39  180.25
   39.68   180.4   40.13   180.5      41  180.64   53.56   182.7   64.04  184.27
   65.91  184.34   68.17  184.59    72.8  184.92   82.01  185.68
#Mann= 3 , 0 , 0
       0    .057       0   37.43     .04       0   39.68    .057       0
Bank Sta=37.43,39.68
XS Rating Curve= 0 ,0
Exp/Cntr=0.3,0.1

Type RM Length L Ch R = 1 ,4727.54 ,19.26,20,19.72
XS GIS Cut Line= 4
342396.6063232425421408.54730225342417.0162963875421413.36407471
342443.3679199225421407.66790771342470.1505126955421385.22271729
#Sta/Elev= 22
       0  186.73    4.63  186.04    6.12  185.87    6.93  185.74   15.09  184.56
   20.97  183.26   24.07  182.65    26.6  181.37   30.23  179.76   32.67  179.74
   34.33  179.65   36.61  179.53   42.07 179.225   44.84  179.02   45.24 179.254
   47.93  180.49   49.08  181.23   53.41  182.09   54.95  182.14    61.7  182.47
   75.76  184.04   82.88  184.57
#Mann= 3 , 0 , 0
       0    .057       0   42.07    .037       0   45.24    .057       0
Bank Sta=42.07,45.24
XS Rating Curve= 0 ,0
Exp/Cntr=0.3,0.1

Type RM Length L Ch R = 1 ,4707.54 ,5.01,5.31,4.99
XS GIS Cut Line= 3
342405.9539184575421428.78527832342427.0795288095421431.20550537
342478.2404785165421415.30487061
#Sta/Elev= 25
       0  184.77      .8  184.65    3.41  184.08   11.15  183.67   15.84  183.34
   16.68  183.26   16.74  183.25   21.26  180.85   21.27  180.85   21.89  180.52
   23.25  179.93   30.32  178.96   33.06  178.28   33.98  178.05   37.37  178.05
    38.6  178.03      40  177.96   42.46 178.064    49.2  178.21    52.4  179.92
   65.34  182.16   67.64  182.47   69.94  182.91   71.52  183.07   74.84  183.28
#Mann= 3 , 0 , 0
       0    .057       0   37.37    .037       0   42.46    .057       0
Bank Sta=37.37,42.46
XS Rating Curve= 0 ,0
Exp/Cntr=0.3,0.1

Type RM Length L Ch R = 1 ,4702.24 ,16.74,19.76,23.42
XS GIS Cut Line= 3
342405.385681152 5421433.7454834342427.5565185555421436.28552246
342479.7224731455421420.07269287
#Sta/Elev= 26
       0  184.64     .14  184.64    6.11  184.07   17.04  183.14   17.44   183.1
   18.41  182.89   22.32  180.69    23.2  180.19   23.51     180   25.32  179.87
   31.43  179.52   32.12  179.47   32.25  179.47   32.66  179.41   33.13  179.29
   36.37  177.95   36.94  177.65   40.39  177.97   41.34  177.99   52.12  178.24
   54.39  179.44   69.79  182.11   72.26  182.82   74.72  182.94   75.35  182.95
   76.94  183.01
#Mann= 3 , 0 , 0
       0    .057       0   36.37    .037       0   40.39    .057       0
Bank Sta=36.37,40.39
XS Rating Curve= 0 ,0
Exp/Cntr=0.3,0.1

Type RM Length L Ch R = 1 ,4682.48 ,24.78,23.69,17.54
XS GIS Cut Line= 3
342384.6652832035421449.13708496342462.1015014655421451.67608643
342490.3955078135421431.71368408
#Sta/Elev= 21
       0  184.23    6.08  183.17    7.27  183.08    27.1  183.85   40.25  182.68
   40.66  182.59   42.69  181.43   45.75  179.52   49.09  179.24   49.65  179.13
   55.24 176.766   55.42  176.63   59.29  176.91   67.95  177.33   77.48   178.4
   83.28  178.87   88.85  180.58   90.14  180.79   92.25   181.5   97.37  181.89
  112.11  182.74
#Mann= 3 , 0 , 0
       0    .057       0   55.24    .037       0   59.29    .057       0
Bank Sta=55.24,59.29
XS Rating Curve= 0 ,0
Exp/Cntr=0.3,0.1

Type RM Length L Ch R = 1 ,4658.79 ,20.47,25.37,24.27
XS GIS Cut Line= 4
342413.6375122075421476.55328369342443.7119140635421474.82592773
 342454.427917485421468.95349121342486.5764770515421446.49951172
#Sta/Elev= 20
       0  183.73   14.57     183   17.96  181.58   23.03  177.93   24.07  177.84
   30.12  176.43   31.78  175.78   32.09  175.59   33.83   175.5    34.4  175.73
   37.22  177.27   38.05  177.54   39.65  177.77   46.28  178.19   50.19  178.31
   57.87  178.75   65.04  179.53    65.9  179.53   69.41  180.72   81.56  181.64
#Mann= 3 , 0 , 0
       0    .057       0   31.78    .037       0    34.4    .057       0
Bank Sta=31.78,34.4
XS Rating Curve= 0 ,0
Exp/Cntr=0.3,0.1

Type RM Length L Ch R = 1 ,4633.41 ,27.81,23.8,18.32
XS GIS Cut Line= 4
342416.7960815435421491.53570557342437.1434936525421493.58789063
342478.5769042975421484.43591309342504.669311523 5421459.3939209
#Sta/Elev= 24
       0  183.21   13.96  182.53   17.01  180.89   20.45  180.15   24.58  178.73
   28.12  177.31   29.03  177.03   29.55  176.87   36.76  176.05   38.89  175.38
   47.43  174.88   49.43  174.77   50.68 174.697   52.47  174.51   52.79  174.66
   53.59  174.98   58.46  177.06    59.2  177.48   62.88  177.18   63.67  177.12
   68.66  177.81   74.47   179.5   84.38  180.18   99.05  181.43
#Mann= 3 , 0 , 0
       0    .057       0   50.68    .037       0   52.79    .057       0
Bank Sta=50.68,52.79
XS Rating Curve= 0 ,0
Exp/Cntr=0.3,0.1
